--- Exploits_FMM.prj (project) ---

Proj Title=Exploits_FMM
Current Plan=p02
Default Exp/Contr=0.3,0.1
SI Units
Geom File=g01
Flow File=f01
Flow File=f02
Plan File=p01
Plan File=p02
Y Axis Title=Elevation
X Axis Title(PF)=Main Channel Distance
X Axis Title(XS)=Station
BEGIN DESCRIPTION:
END DESCRIPTION:
DSS Export Rating Curves= 0
DSS Export Rating Curve Sorted= 0
DSS Export Volume Flow Curves= 0
DXF OffsetX= 0
DXF OffsetY= 0
DXF ScaleX= 1
DXF ScaleY= 10

--- Exploits_FMM.p02 (plan) ---

Plan Title=2021_05_13_GF_Mods
Program Version=5.06
Short Identifier=2021_05_13
Geom File=g01
Flow File=f02
Mixed Flow
K Sum by GR= 0
Std Step Tol= 0.003
Critical Tol= 0.003
Num of Std Step Trials= 20
Max Error Tol= 0.1
Flow Tol Ratio= 0.001
Split Flow NTrial= 30
Split Flow Tol= 0.006
Split Flow Ratio= 0.02
Log Output Level= 0
Friction Slope Method= 1
Unsteady Friction Slope Method= 2
Unsteady Bridges Friction Slope Method= 1
Parabolic Critical Depth
Global Vel Dist= 0 , 0 , 0
Global Log Level= 0
CheckData=True
Encroach Param=-1 ,0,0, 0
Optimized Weir=Exploits River  ,CB to BF4       ,43.309
Optimized Weir=Exploits River  ,CB to BF4       ,43.231
BEGIN DESCRIPTION:
Plan for "Exploits" runs (1:20 CC - Exploits, 1:20 CLC - Exploits, 1:100 CC - Exploits, 1:100 CLC Exploits)
Properly represents flow split between GF Main Dam and GF Power Canal in Exploits runs.
END DESCRIPTION:
Computation Interval=1MIN
Output Interval=1HOUR
Instantaneous Interval=1HOUR
Mapping Interval=1HOUR
Computation Time Step Use Courant=        0
Computation Time Step Use Time Series=    0
Computation Time Step Count To Double=0
Computation Time Step Max Doubling=0
Computation Time Step Max Halving=0
Computation Time Step Residence Courant=0
Run HTab= 0
Run UNet= 0
Run Sediment= 0
Run PostProcess= 0
Run WQNet= 0
Run RASMapper= 0
UNET Theta= 1
UNET Theta Warmup= 1
UNET ZTol= 0.006
UNET ZSATol= 0.006
UNET MxIter= 20
UNET Max Iter WO Improvement= 0
UNET MaxInSteps= 0
UNET DtIC= 0
UNET DtMin= 0
UNET MaxCRTS= 20
UNET WFStab= 2
UNET SFStab= 1
UNET WFX= 1
UNET SFX= 1
UNET 1D Methodology=Finite Difference
UNET DSS MLevel= 4
UNET Pardiso=0
UNET DZMax Abort= 30
UNET Use Existing IB Tables=-1
UNET Froude Reduction=False
UNET Froude Limit= 0.8
UNET Froude Power= 4
UNET D1 Cores= 0
UNET D2 Coriolis=0
UNET D2 Cores= 0
UNET D2 Theta= 1
UNET D2 Theta Warmup= 1
UNET D2 Z Tol= 0.003
UNET D2 Volume Tol= 0.003
UNET D2 Max Iterations= 20
UNET D2 Equation= 0
UNET D2 RampUpFraction=0.1
UNET D2 TimeSlices= 1
UNET D2 BCVolumeCheck=0
UNET D1D2 MaxIter= 0
UNET D1D2 ZTol=0.003
UNET D1D2 QTol=0.1
UNET D1D2 MinQTol=0.03
Write IC File= 0
Write IC File at Fixed DateTime=0
Write IC File at Sim End=0
Echo Input=False
Echo Parameters=False
Echo Output=False
Write Detailed= 0
HDF Write Warmup=0
HDF Write Time Slices=0
HDF Flush=0
HDF Face Node Velocities=0
HDF Compression= 1
HDF Chunk Size= 1
HDF Spatial Parts= 1
HDF Use Max Rows=0
HDF Fixed Rows= 1
Calibration Method= 0
Calibration Iterations= 20
Calibration Max Change=0.05
Calibration Tolerance=0.2
Calibration Maximum=1.5
Calibration Minimum=0.5
Calibration Optimization Method= 1
WQ AD Non Conservative
WQ ULTIMATE=-1
WQ Max Comp Step=1HOUR
WQ Output Interval=15MIN
WQ Output Selected Increments= 0
WQ Output face flow=0
WQ Output face velocity=0
WQ Output face area=0
WQ Output face dispersion=0
WQ Output cell volume=0
WQ Output cell surface area=0
WQ Output cell continuity=0
WQ Output cumulative cell continuity=0
WQ Output face conc=0
WQ Output face dconc_dx=0
WQ Output face courant=0
WQ Output face peclet=0
WQ Output face adv mass=0
WQ Output face disp mass=0
WQ Output cell mass=0
WQ Output cell source sink temp=0
WQ Output nsm pathways=0
WQ Output nsm derived pathways=0
WQ Output MaxMinRange=-1
WQ Daily Max Min Mean=-1
WQ Daily Range=0
WQ Daily Time=0
WQ Create Restart=0
WQ Fixed Restart=0
WQ System Summary=0
WQ Write To DSS=0
WQ Use Fixed Temperature=0
Sorting and Armoring Iterations= 10
XS Update Threshold= 0.02
Bed Roughness Predictor= 0
Hydraulics Update Threshold= 0.02
Energy Slope Method= 1
Volume Change Method= 1
Sediment Retention Method= 0
XS Weighting Method= 0
Number of US Weighted Cross Sections= 1
Number of DS Weighted Cross Sections= 1
Upstream XS Weight=0
Main XS Weight=1
Downstream XS Weight=0
Number of DS XS's Weighted with US Boundary= 1
Upstream Boundary Weight= 1
Weight of XSs Associated with US Boundary= 0
Number of US XS's Weighted with DS Boundary= 1
Downstream Boundary Weight= 0.5
Weight of XSs Associated with DS Boundary= 0.5
Percentile Method= 0
Sediment Output Level= 3
Mass or Volume Output= 0
Output Increment Type= 1
Profile and TS Output Increment= 1
XS Output Flag= 0
XS Output Increment= 10
Write Gradation File= 0
Read Gradation Hotstart= 0
Write HDF5 File= 1
Write Binary Output= 1
Write DSS Sediment File= 0
SV Curve= 0
Specific Gage Flag= 0

--- Exploits_FMM.p01 (plan) ---

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Plan Title=2021_02_09
Short Identifier=2021Feb09
Geom File=g01
Flow File=f01
Plan for "Tributary" runs (1:20 CC - Tribs, 1:20 CLC - Tribs, 1:100 CC - Tribs, 1:100 CLC Tribs)

--- Exploits_FMM.f02 (steady flow) ---

Flow Title=2021_05_13_SteadyFlows_GF_Mods
Program Version=5.06
BEGIN FILE DESCRIPTION:
Adjusted elevation of Grand Falls Power Canal to properly represent flow split between GF Main Dam and GF Power Canal in Exploits runs.
END FILE DESCRIPTION:
Number of Profiles= 8
Profile Names=1:20 CC - Exploits,1:20 CLC - Exploits,1:100 CC - Exploits,1:100 CLC - Exploits,1:20 CC - Tribs,1:20 CLC - Tribs,1:100 CC - Tribs,1:100 CLC - Tribs
River Rch & RM=B1,B1              ,0.9685
     .01     .01     .01     .01     5.4     6.4       7     8.1
River Rch & RM=Badger Brk,Badger Brk      ,1.9217
     .01     .01     .01     .01     257281.0938     325344.2635
River Rch & RM=BF1,BF1             ,1.2199
     .01     .01     .01     .01     .01     .01     .01     .01
River Rch & RM=BF1,BF1             ,.3504
     .01     .01     .01     .01      .3      .3      .4      .4
River Rch & RM=BF2,BF2             ,1.2490
     .01     .01     .01     .013.0143543.5669863.8684214.471292
River Rch & RM=BF2,BF2             ,0.8133
     .01     .01     .01     .014.8229675.7071776.1894747.154067
River Rch & RM=BF3,BF3             ,2.1832
     .01     .01     .01     .01     7.6     8.5      10      11
River Rch & RM=BF3,BF3             ,0.8646
     .01     .01     .01     .01     7.6     8.6    10.2    11.2
River Rch & RM=BF4,BF4             ,0.9422
     .01     .01     .01     .011.0942281.2563361.3779171.580552
River Rch & RM=BF4,BF4             ,0.6155
     .01     .01     .01     .011.4014931.6091221.7648432.024379
River Rch & RM=Corduroy Brk,Corduroy Brk    ,3.8918
     .01     .01     .01     .01     4.6       5     5.6     6.3
River Rch & RM=Corduroy Brk,Corduroy Brk    ,3.2308
     .01     .01     .01     .01     3.6     3.6     3.6     3.6
River Rch & RM=Corduroy Brk,Corduroy Brk    ,2.5346
     .01     .01     .01     .01       4     4.3     4.9     5.6
River Rch & RM=Corduroy Brk,Corduroy Brk    ,1.7767
     .01     .01     .01     .01     6.1     6.7     7.2     8.1
River Rch & RM=Corduroy Brk,Corduroy Brk    ,1.3922
     .01     .01     .01     .01       7     7.4     7.8     8.2
River Rch & RM=Corduroy Brk,Corduroy Brk    ,0.7838
     .01     .01     .01     .01    10.2    10.9    11.5    12.3
River Rch & RM=Exploits River,Mill to LRI     ,127.9419
    13401468.405    16501747.339     .01     .01     .01     .01
River Rch & RM=Exploits River,Mill to LRI     ,98.9083
    13401468.405    16501747.339     .01     .01     .01     .01
River Rch & RM=Exploits River,LRI to Badger   ,75.6731
    14001535.016    1715 1816.68     .01     .01     .01     .01
River Rch & RM=Exploits River,Badger to Wigwam,75.2189
    14181553.786    17301832.852     .01     .01     .01     .01
River Rch & RM=Exploits River,Badger to Wigwam,54.2773
    14301563.804    1740 1839.12     .01     .01     .01     .01
River Rch & RM=Exploits River,Wigwam to RP    ,49.8124
    14301563.804    1740 1839.12     .01     .01     .01     .01
River Rch & RM=Exploits River,RP to CB        ,48.3493
    14301563.804    1740 1839.12     .01     .01     .01     .01
River Rch & RM=Exploits River,RP to CB        ,46.8155
    14981638.733    18181922.646     .01     .01     .01     .01
River Rch & RM=Exploits River,CB to BF4       ,43.6571
    14981638.733    18181922.646     .01     .01     .01     .01
River Rch & RM=Exploits River,CB to BF4       ,43.2587
    15001641.405    18201924.198     .01     .01     .01     .01
River Rch & RM=Exploits River,BF4 to BF3      ,28.6539
    15001641.405    18201924.198     .01     .01     .01     .01
River Rch & RM=Exploits River,BF3 to BF2      ,25.6408
    15001641.405    18201924.198     .01     .01     .01     .01
River Rch & RM=Exploits River,BF3 to BF2      ,23.7672
    22202435.927    28102975.312     .01     .01     .01     .01
River Rch & RM=Exploits River,BF2 to BF1      ,23.3904
    22202435.927    28102975.312     .01     .01     .01     .01
River Rch & RM=Exploits River,BF1 to Outlet   ,20.2457
    22202435.927    28102975.312     .01     .01     .01     .01
River Rch & RM=GF1,GF1             ,3.9291
     .01     .01     .01     .01       1     1.2     1.3     1.5
River Rch & RM=GF1,GF1             ,3.1868
     .01     .01     .01     .01     1.5   1.775   1.925    2.25
River Rch & RM=GF1,GF1             ,1.9833
     .01     .01     .01     .01       6     7.1     7.7       9
River Rch & RM=GF1,GF1             ,1.0726
     .01     .01     .01     .01    13.9    15.9    17.9      20
River Rch & RM=Little Red Ind,LRI to B1       ,1.4448
     .01     .01     .01     .01    77.5 85.4754     101107.5051
River Rch & RM=Little Red Ind,B1 to Expl      ,1.2620
     .01     .01     .01     .01    82.991.87539     108115.6051
River Rch & RM=Little Rushy Pd,Little Rushy Pd ,0.5608
     .01     .01     .01     .01     1.9     2.1     2.4     2.7
River Rch & RM=Mullens Pond,Mullens Pond    ,0.4097
     .01     .01     .01     .01     1.7       2     2.1     2.5
River Rch & RM=Rushy Pond,Rushy Pond      ,1.605
     .01     .01     .01     .01    22.8    25.7    29.6    32.7
River Rch & RM=Wigwam Brook,Wigwam Brook    ,4.6443
     .01     .01     .01     .01    18.8    21.3    24.4      27
River Rch & RM=Wigwam Brook,Wigwam Brook    ,3.5404
     .01     .01     .01     .01    26.2    29.8    33.9    37.8
Boundary for River Rch & Prof#=B1,B1              , 1
Up Type= 3
Up Slope=1.911504E-03
Dn Type= 0
Boundary for River Rch & Prof#=B1,B1              , 2
Up Type= 3
Up Slope=1.911504E-03
Dn Type= 0
Boundary for River Rch & Prof#=B1,B1              , 3
Up Type= 3
Up Slope=1.911504E-03
Dn Type= 0
Boundary for River Rch & Prof#=B1,B1              , 4
Up Type= 3
Up Slope=1.911504E-03
Dn Type= 0
Boundary for River Rch & Prof#=B1,B1              , 5
Up Type= 3
Up Slope=1.911504E-03
Dn Type= 0
Boundary for River Rch & Prof#=B1,B1              , 6
Up Type= 3
Up Slope=1.911504E-03
Dn Type= 0
Boundary for River Rch & Prof#=B1,B1              , 7
Up Type= 3
Up Slope=1.911504E-03
Dn Type= 0
Boundary for River Rch & Prof#=B1,B1              , 8
Up Type= 3
Up Slope=1.911504E-03
Dn Type= 0
Boundary for River Rch & Prof#=Badger Brk,Badger Brk      , 1
Up Type= 3
Up Slope=0.00004
Dn Type= 0
Boundary for River Rch & Prof#=Badger Brk,Badger Brk      , 2
Up Type= 3
Up Slope=0.00004
Dn Type= 0
Boundary for River Rch & Prof#=Badger Brk,Badger Brk      , 3
Up Type= 3
Up Slope=0.00004
Dn Type= 0
Boundary for River Rch & Prof#=Badger Brk,Badger Brk      , 4
Up Type= 3
Up Slope=0.00004
Dn Type= 0
Boundary for River Rch & Prof#=Badger Brk,Badger Brk      , 5
Up Type= 3
Up Slope=0.00004
Dn Type= 0
Boundary for River Rch & Prof#=Badger Brk,Badger Brk      , 6
Up Type= 3
Up Slope=0.00004
Dn Type= 0
Boundary for River Rch & Prof#=Badger Brk,Badger Brk      , 7
Up Type= 3
Up Slope=0.00004
Dn Type= 0
Boundary for River Rch & Prof#=Badger Brk,Badger Brk      , 8
Up Type= 3
Up Slope=0.00004
Dn Type= 0
Boundary for River Rch & Prof#=BF1,BF1             , 1
Up Type= 3
Up Slope=5.857143E-03
Dn Type= 0
Boundary for River Rch & Prof#=BF1,BF1             , 2
Up Type= 3
Up Slope=5.857143E-03
Dn Type= 0
Boundary for River Rch & Prof#=BF1,BF1             , 3
Up Type= 3
Up Slope=5.857143E-03
Dn Type= 0
Boundary for River Rch & Prof#=BF1,BF1             , 4
Up Type= 3
Up Slope=5.857143E-03
Dn Type= 0
Boundary for River Rch & Prof#=BF1,BF1             , 5
Up Type= 3
Up Slope=5.857143E-03
Dn Type= 0
Boundary for River Rch & Prof#=BF1,BF1             , 6
Up Type= 3
Up Slope=5.857143E-03
Dn Type= 0
Boundary for River Rch & Prof#=BF1,BF1             , 7
Up Type= 3
Up Slope=5.857143E-03
Dn Type= 0
Boundary for River Rch & Prof#=BF1,BF1             , 8
Up Type= 3
Up Slope=5.857143E-03
Dn Type= 0
Boundary for River Rch & Prof#=BF2,BF2             , 1
Up Type= 3
Up Slope=1.396614E-02
Dn Type= 0
Boundary for River Rch & Prof#=BF2,BF2             , 2
Up Type= 3
Up Slope=1.396614E-02
Dn Type= 0
Boundary for River Rch & Prof#=BF2,BF2             , 3
Up Type= 3
Up Slope=1.396614E-02
Dn Type= 0
Boundary for River Rch & Prof#=BF2,BF2             , 4
Up Type= 3
Up Slope=1.396614E-02
Dn Type= 0
Boundary for River Rch & Prof#=BF2,BF2             , 5
Up Type= 3
Up Slope=1.396614E-02
Dn Type= 0
Boundary for River Rch & Prof#=BF2,BF2             , 6
Up Type= 3
Up Slope=1.396614E-02
Dn Type= 0
Boundary for River Rch & Prof#=BF2,BF2             , 7
Up Type= 3
Up Slope=1.396614E-02
Dn Type= 0
Boundary for River Rch & Prof#=BF2,BF2             , 8
Up Type= 3
Up Slope=1.396614E-02
Dn Type= 0
Boundary for River Rch & Prof#=BF3,BF3             , 1
Up Type= 3
Up Slope=2.193798E-03
Dn Type= 0
Boundary for River Rch & Prof#=BF3,BF3             , 2
Up Type= 3
Up Slope=2.193798E-03
Dn Type= 0
Boundary for River Rch & Prof#=BF3,BF3             , 3
Up Type= 3
Up Slope=2.193798E-03
Dn Type= 0
Boundary for River Rch & Prof#=BF3,BF3             , 4
Up Type= 3
Up Slope=2.193798E-03
Dn Type= 0
Boundary for River Rch & Prof#=BF3,BF3             , 5
Up Type= 3
Up Slope=2.193798E-03
Dn Type= 0
Boundary for River Rch & Prof#=BF3,BF3             , 6
Up Type= 3
Up Slope=2.193798E-03
Dn Type= 0
Boundary for River Rch & Prof#=BF3,BF3             , 7
Up Type= 3
Up Slope=2.193798E-03
Dn Type= 0
Boundary for River Rch & Prof#=BF3,BF3             , 8
Up Type= 3
Up Slope=2.193798E-03
Dn Type= 0
Boundary for River Rch & Prof#=BF4,BF4             , 1
Up Type= 3
Up Slope=4.040541E-03
Dn Type= 0
Boundary for River Rch & Prof#=BF4,BF4             , 2
Up Type= 3
Up Slope=4.040541E-03
Dn Type= 0
Boundary for River Rch & Prof#=BF4,BF4             , 3
Up Type= 3
Up Slope=4.040541E-03
Dn Type= 0
Boundary for River Rch & Prof#=BF4,BF4             , 4
Up Type= 3
Up Slope=4.040541E-03
Dn Type= 0
Boundary for River Rch & Prof#=BF4,BF4             , 5
Up Type= 3
Up Slope=4.040541E-03
Dn Type= 0
Boundary for River Rch & Prof#=BF4,BF4             , 6
Up Type= 3
Up Slope=4.040541E-03
Dn Type= 0
Boundary for River Rch & Prof#=BF4,BF4             , 7
Up Type= 3
Up Slope=4.040541E-03
Dn Type= 0
Boundary for River Rch & Prof#=BF4,BF4             , 8
Up Type= 3
Up Slope=4.040541E-03
Dn Type= 0
Boundary for River Rch & Prof#=Corduroy Brk,Corduroy Brk    , 1
Up Type= 3
Up Slope=3.948357E-03
Dn Type= 0
Boundary for River Rch & Prof#=Corduroy Brk,Corduroy Brk    , 2
Up Type= 3
Up Slope=3.948357E-03
Dn Type= 0
Boundary for River Rch & Prof#=Corduroy Brk,Corduroy Brk    , 3
Up Type= 3
Up Slope=3.948357E-03
Dn Type= 0
Boundary for River Rch & Prof#=Corduroy Brk,Corduroy Brk    , 4
Up Type= 3
Up Slope=3.948357E-03
Dn Type= 0
Boundary for River Rch & Prof#=Corduroy Brk,Corduroy Brk    , 5
Up Type= 3
Up Slope=3.948357E-03
Dn Type= 0
Boundary for River Rch & Prof#=Corduroy Brk,Corduroy Brk    , 6
Up Type= 3
Up Slope=3.948357E-03
Dn Type= 0
Boundary for River Rch & Prof#=Corduroy Brk,Corduroy Brk    , 7
Up Type= 3
Up Slope=3.948357E-03
Dn Type= 0
Boundary for River Rch & Prof#=Corduroy Brk,Corduroy Brk    , 8
Up Type= 3
Up Slope=3.948357E-03
Dn Type= 0
Boundary for River Rch & Prof#=Exploits River,Mill to LRI     , 1
Up Type= 1
Up Known WS=146.6381
Dn Type= 0
Boundary for River Rch & Prof#=Exploits River,Mill to LRI     , 2
Up Type= 1
Up Known WS=146.6381
Dn Type= 0
Boundary for River Rch & Prof#=Exploits River,Mill to LRI     , 3
Up Type= 1
Up Known WS=146.6381
Dn Type= 0
Boundary for River Rch & Prof#=Exploits River,Mill to LRI     , 4
Up Type= 1
Up Known WS=146.6381
Dn Type= 0
Boundary for River Rch & Prof#=Exploits River,Mill to LRI     , 5
Up Type= 1
Up Known WS=146.6381
Dn Type= 0
Boundary for River Rch & Prof#=Exploits River,Mill to LRI     , 6
Up Type= 1
Up Known WS=146.6381
Dn Type= 0
Boundary for River Rch & Prof#=Exploits River,Mill to LRI     , 7
Up Type= 1
Up Known WS=146.6381
Dn Type= 0
Boundary for River Rch & Prof#=Exploits River,Mill to LRI     , 8
Up Type= 1
Up Known WS=146.6381
Dn Type= 0
Boundary for River Rch & Prof#=Exploits River,LRI to Badger   , 1
Up Type= 0
Dn Type= 0
Boundary for River Rch & Prof#=Exploits River,LRI to Badger   , 2
Up Type= 0
Dn Type= 0
Boundary for River Rch & Prof#=Exploits River,LRI to Badger   , 3
Up Type= 0
Dn Type= 0
Boundary for River Rch & Prof#=Exploits River,LRI to Badger   , 4
Up Type= 0
Dn Type= 0
Boundary for River Rch & Prof#=Exploits River,LRI to Badger   , 5
Up Type= 0
Dn Type= 0
Boundary for River Rch & Prof#=Exploits River,LRI to Badger   , 6
Up Type= 0
Dn Type= 0
Boundary for River Rch & Prof#=Exploits River,LRI to Badger   , 7
Up Type= 0
Dn Type= 0
Boundary for River Rch & Prof#=Exploits River,LRI to Badger   , 8
Up Type= 0
Dn Type= 0
Boundary for River Rch & Prof#=Exploits River,Badger to Wigwam, 1
Up Type= 0
Dn Type= 0
Boundary for River Rch & Prof#=Exploits River,Badger to Wigwam, 2
Up Type= 0
Dn Type= 0
Boundary for River Rch & Prof#=Exploits River,Badger to Wigwam, 3
Up Type= 0
Dn Type= 0
Boundary for River Rch & Prof#=Exploits River,Badger to Wigwam, 4
Up Type= 0
Dn Type= 0
Boundary for River Rch & Prof#=Exploits River,Badger to Wigwam, 5
Up Type= 0
Dn Type= 0
Boundary for River Rch & Prof#=Exploits River,Badger to Wigwam, 6
Up Type= 0
Dn Type= 0
Boundary for River Rch & Prof#=Exploits River,Badger to Wigwam, 7
Up Type= 0
Dn Type= 0
Boundary for River Rch & Prof#=Exploits River,Badger to Wigwam, 8
Up Type= 0
Dn Type= 0
Boundary for River Rch & Prof#=Exploits River,Wigwam to RP    , 1
Up Type= 0
Dn Type= 0
Boundary for River Rch & Prof#=Exploits River,Wigwam to RP    , 2
Up Type= 0
Dn Type= 0
Boundary for River Rch & Prof#=Exploits River,Wigwam to RP    , 3
Up Type= 0
Dn Type= 0
Boundary for River Rch & Prof#=Exploits River,Wigwam to RP    , 4
Up Type= 0
Dn Type= 0
Boundary for River Rch & Prof#=Exploits River,Wigwam to RP    , 5
Up Type= 0
Dn Type= 0
Boundary for River Rch & Prof#=Exploits River,Wigwam to RP    , 6
Up Type= 0
Dn Type= 0
Boundary for River Rch & Prof#=Exploits River,Wigwam to RP    , 7
Up Type= 0
Dn Type= 0
Boundary for River Rch & Prof#=Exploits River,Wigwam to RP    , 8
Up Type= 0
Dn Type= 0
Boundary for River Rch & Prof#=Exploits River,RP to CB        , 1
Up Type= 0
Dn Type= 0
Boundary for River Rch & Prof#=Exploits River,RP to CB        , 2
Up Type= 0
Dn Type= 0
Boundary for River Rch & Prof#=Exploits River,RP to CB        , 3
Up Type= 0
Dn Type= 0
Boundary for River Rch & Prof#=Exploits River,RP to CB        , 4
Up Type= 0
Dn Type= 0
Boundary for River Rch & Prof#=Exploits River,RP to CB        , 5
Up Type= 0
Dn Type= 0
Boundary for River Rch & Prof#=Exploits River,RP to CB        , 6
Up Type= 0
Dn Type= 0
Boundary for River Rch & Prof#=Exploits River,RP to CB        , 7
Up Type= 0
Dn Type= 0
Boundary for River Rch & Prof#=Exploits River,RP to CB        , 8
Up Type= 0
Dn Type= 0
Boundary for River Rch & Prof#=Exploits River,CB to BF4       , 1
Up Type= 0
Dn Type= 0
Boundary for River Rch & Prof#=Exploits River,CB to BF4       , 2
Up Type= 0
Dn Type= 0
Boundary for River Rch & Prof#=Exploits River,CB to BF4       , 3
Up Type= 0
Dn Type= 0
Boundary for River Rch & Prof#=Exploits River,CB to BF4       , 4
Up Type= 0
Dn Type= 0
Boundary for River Rch & Prof#=Exploits River,CB to BF4       , 5
Up Type= 0
Dn Type= 0
Boundary for River Rch & Prof#=Exploits River,CB to BF4       , 6
Up Type= 0
Dn Type= 0
Boundary for River Rch & Prof#=Exploits River,CB to BF4       , 7
Up Type= 0
Dn Type= 0
Boundary for River Rch & Prof#=Exploits River,CB to BF4       , 8
Up Type= 0
Dn Type= 0
Boundary for River Rch & Prof#=Exploits River,BF4 to BF3      , 1
Up Type= 0
Dn Type= 0
Boundary for River Rch & Prof#=Exploits River,BF4 to BF3      , 2
Up Type= 0
Dn Type= 0
Boundary for River Rch & Prof#=Exploits River,BF4 to BF3      , 3
Up Type= 0
Dn Type= 0
Boundary for River Rch & Prof#=Exploits River,BF4 to BF3      , 4
Up Type= 0
Dn Type= 0
Boundary for River Rch & Prof#=Exploits River,BF4 to BF3      , 5
Up Type= 0
Dn Type= 0
Boundary for River Rch & Prof#=Exploits River,BF4 to BF3      , 6
Up Type= 0
Dn Type= 0
Boundary for River Rch & Prof#=Exploits River,BF4 to BF3      , 7
Up Type= 0
Dn Type= 0
Boundary for River Rch & Prof#=Exploits River,BF4 to BF3      , 8
Up Type= 0
Dn Type= 0
Boundary for River Rch & Prof#=Exploits River,BF3 to BF2      , 1
Up Type= 0
Dn Type= 0
Boundary for River Rch & Prof#=Exploits River,BF3 to BF2      , 2
Up Type= 0
Dn Type= 0
Boundary for River Rch & Prof#=Exploits River,BF3 to BF2      , 3
Up Type= 0
Dn Type= 0
Boundary for River Rch & Prof#=Exploits River,BF3 to BF2      , 4
Up Type= 0
Dn Type= 0
Boundary for River Rch & Prof#=Exploits River,BF3 to BF2      , 5
Up Type= 0
Dn Type= 0
Boundary for River Rch & Prof#=Exploits River,BF3 to BF2      , 6
Up Type= 0
Dn Type= 0
Boundary for River Rch & Prof#=Exploits River,BF3 to BF2      , 7
Up Type= 0
Dn Type= 0
Boundary for River Rch & Prof#=Exploits River,BF3 to BF2      , 8
Up Type= 0
Dn Type= 0
Boundary for River Rch & Prof#=Exploits River,BF2 to BF1      , 1
Up Type= 0
Dn Type= 0
Boundary for River Rch & Prof#=Exploits River,BF2 to BF1      , 2
Up Type= 0
Dn Type= 0
Boundary for River Rch & Prof#=Exploits River,BF2 to BF1      , 3
Up Type= 0
Dn Type= 0
Boundary for River Rch & Prof#=Exploits River,BF2 to BF1      , 4
Up Type= 0
Dn Type= 0
Boundary for River Rch & Prof#=Exploits River,BF2 to BF1      , 5
Up Type= 0
Dn Type= 0
Boundary for River Rch & Prof#=Exploits River,BF2 to BF1      , 6
Up Type= 0
Dn Type= 0
Boundary for River Rch & Prof#=Exploits River,BF2 to BF1      , 7
Up Type= 0
Dn Type= 0
Boundary for River Rch & Prof#=Exploits River,BF2 to BF1      , 8
Up Type= 0
Dn Type= 0
Boundary for River Rch & Prof#=Exploits River,BF1 to Outlet   , 1
Up Type= 0
Dn Type= 1
Dn Known WS=0.4
Boundary for River Rch & Prof#=Exploits River,BF1 to Outlet   , 2
Up Type= 0
Dn Type= 1
Dn Known WS=1.3
Boundary for River Rch & Prof#=Exploits River,BF1 to Outlet   , 3
Up Type= 0
Dn Type= 1
Dn Known WS=0.4
Boundary for River Rch & Prof#=Exploits River,BF1 to Outlet   , 4
Up Type= 0
Dn Type= 1
Dn Known WS=1.3
Boundary for River Rch & Prof#=Exploits River,BF1 to Outlet   , 5
Up Type= 0
Dn Type= 1
Dn Known WS=0.4
Boundary for River Rch & Prof#=Exploits River,BF1 to Outlet   , 6
Up Type= 0
Dn Type= 1
Dn Known WS=0.4
Boundary for River Rch & Prof#=Exploits River,BF1 to Outlet   , 7
Up Type= 0
Dn Type= 1
Dn Known WS=0.4
Boundary for River Rch & Prof#=Exploits River,BF1 to Outlet   , 8
Up Type= 0
Dn Type= 1
Dn Known WS=0.4
Boundary for River Rch & Prof#=GF1,GF1             , 1
Up Type= 3
Up Slope=0.0180531
Dn Type= 3
Dn Slope=2.026667E-02
Boundary for River Rch & Prof#=GF1,GF1             , 2
Up Type= 3
Up Slope=0.0180531
Dn Type= 3
Dn Slope=2.026667E-02
Boundary for River Rch & Prof#=GF1,GF1             , 3
Up Type= 3
Up Slope=0.0180531
Dn Type= 3
Dn Slope=2.026667E-02
Boundary for River Rch & Prof#=GF1,GF1             , 4
Up Type= 3
Up Slope=0.0180531
Dn Type= 3
Dn Slope=2.026667E-02
Boundary for River Rch & Prof#=GF1,GF1             , 5
Up Type= 3
Up Slope=0.0180531
Dn Type= 3
Dn Slope=2.026667E-02
Boundary for River Rch & Prof#=GF1,GF1             , 6
Up Type= 3
Up Slope=0.0180531
Dn Type= 3
Dn Slope=2.026667E-02
Boundary for River Rch & Prof#=GF1,GF1             , 7
Up Type= 3
Up Slope=0.0180531
Dn Type= 3
Dn Slope=2.026667E-02
Boundary for River Rch & Prof#=GF1,GF1             , 8
Up Type= 3
Up Slope=0.0180531
Dn Type= 3
Dn Slope=2.026667E-02
Boundary for River Rch & Prof#=Little Red Ind,LRI to B1       , 1
Up Type= 3
Up Slope=0.001464
Dn Type= 0
Boundary for River Rch & Prof#=Little Red Ind,LRI to B1       , 2
Up Type= 3
Up Slope=0.001464
Dn Type= 0
Boundary for River Rch & Prof#=Little Red Ind,LRI to B1       , 3
Up Type= 3
Up Slope=0.001464
Dn Type= 0
Boundary for River Rch & Prof#=Little Red Ind,LRI to B1       , 4
Up Type= 3
Up Slope=0.001464
Dn Type= 0
Boundary for River Rch & Prof#=Little Red Ind,LRI to B1       , 5
Up Type= 3
Up Slope=0.001464
Dn Type= 0
Boundary for River Rch & Prof#=Little Red Ind,LRI to B1       , 6
Up Type= 3
Up Slope=0.001464
Dn Type= 0
Boundary for River Rch & Prof#=Little Red Ind,LRI to B1       , 7
Up Type= 3
Up Slope=0.001464
Dn Type= 0
Boundary for River Rch & Prof#=Little Red Ind,LRI to B1       , 8
Up Type= 3
Up Slope=0.001464
Dn Type= 0
Boundary for River Rch & Prof#=Little Red Ind,B1 to Expl      , 1
Up Type= 0
Dn Type= 0
Boundary for River Rch & Prof#=Little Red Ind,B1 to Expl      , 2
Up Type= 0
Dn Type= 0
Boundary for River Rch & Prof#=Little Red Ind,B1 to Expl      , 3
Up Type= 0
Dn Type= 0
Boundary for River Rch & Prof#=Little Red Ind,B1 to Expl      , 4
Up Type= 0
Dn Type= 0
Boundary for River Rch & Prof#=Little Red Ind,B1 to Expl      , 5
Up Type= 0
Dn Type= 0
Boundary for River Rch & Prof#=Little Red Ind,B1 to Expl      , 6
Up Type= 0
Dn Type= 0
Boundary for River Rch & Prof#=Little Red Ind,B1 to Expl      , 7
Up Type= 0
Dn Type= 0
Boundary for River Rch & Prof#=Little Red Ind,B1 to Expl      , 8
Up Type= 0
Dn Type= 0
Boundary for River Rch & Prof#=Little Rushy Pd,Little Rushy Pd , 1
Up Type= 3
Up Slope=4.474684E-03
Dn Type= 0
Boundary for River Rch & Prof#=Little Rushy Pd,Little Rushy Pd , 2
Up Type= 3
Up Slope=4.474684E-03
Dn Type= 0
Boundary for River Rch & Prof#=Little Rushy Pd,Little Rushy Pd , 3
Up Type= 3
Up Slope=4.474684E-03
Dn Type= 0
Boundary for River Rch & Prof#=Little Rushy Pd,Little Rushy Pd , 4
Up Type= 3
Up Slope=4.474684E-03
Dn Type= 0
Boundary for River Rch & Prof#=Little Rushy Pd,Little Rushy Pd , 5
Up Type= 3
Up Slope=4.474684E-03
Dn Type= 0
Boundary for River Rch & Prof#=Little Rushy Pd,Little Rushy Pd , 6
Up Type= 3
Up Slope=4.474684E-03
Dn Type= 0
Boundary for River Rch & Prof#=Little Rushy Pd,Little Rushy Pd , 7
Up Type= 3
Up Slope=4.474684E-03
Dn Type= 0
Boundary for River Rch & Prof#=Little Rushy Pd,Little Rushy Pd , 8
Up Type= 3
Up Slope=4.474684E-03
Dn Type= 0
Boundary for River Rch & Prof#=Mullens Pond,Mullens Pond    , 1
Up Type= 3
Up Slope=2.605769E-03
Dn Type= 4
Dn Rating Curve # Pts= 21
       0    72.7      .2   73.15      .4   73.37      .6   73.56      .8   73.74
       1    73.9     1.2   73.95     1.4   73.99     1.6   74.01     1.8   74.03
       2   74.04     2.2   74.06     2.4   74.07     2.6   74.08     2.8   74.09
       3    74.1     3.2    74.1     3.4   74.11     3.6   74.12     3.8   74.12
       4   74.13
Boundary for River Rch & Prof#=Mullens Pond,Mullens Pond    , 2
Up Type= 3
Up Slope=2.605769E-03
Dn Type= 3
Dn Slope=0.02
Boundary for River Rch & Prof#=Mullens Pond,Mullens Pond    , 3
Up Type= 3
Up Slope=2.605769E-03
Dn Type= 3
Dn Slope=0.02
Boundary for River Rch & Prof#=Mullens Pond,Mullens Pond    , 4
Up Type= 3
Up Slope=2.605769E-03
Dn Type= 3
Dn Slope=0.02
Boundary for River Rch & Prof#=Mullens Pond,Mullens Pond    , 5
Up Type= 3
Up Slope=2.605769E-03
Dn Type= 3
Dn Slope=0.02
Boundary for River Rch & Prof#=Mullens Pond,Mullens Pond    , 6
Up Type= 3
Up Slope=2.605769E-03
Dn Type= 3
Dn Slope=0.02
Boundary for River Rch & Prof#=Mullens Pond,Mullens Pond    , 7
Up Type= 3
Up Slope=2.605769E-03
Dn Type= 3
Dn Slope=0.02
Boundary for River Rch & Prof#=Mullens Pond,Mullens Pond    , 8
Up Type= 3
Up Slope=2.605769E-03
Dn Type= 3
Dn Slope=0.02
Boundary for River Rch & Prof#=Rushy Pond,Rushy Pond      , 1
Up Type= 0
Dn Type= 0
Boundary for River Rch & Prof#=Rushy Pond,Rushy Pond      , 2
Up Type= 0
Dn Type= 0
Boundary for River Rch & Prof#=Rushy Pond,Rushy Pond      , 3
Up Type= 0
Dn Type= 0
Boundary for River Rch & Prof#=Rushy Pond,Rushy Pond      , 4
Up Type= 0
Dn Type= 0
Boundary for River Rch & Prof#=Rushy Pond,Rushy Pond      , 5
Up Type= 0
Dn Type= 0
Boundary for River Rch & Prof#=Rushy Pond,Rushy Pond      , 6
Up Type= 0
Dn Type= 0
Boundary for River Rch & Prof#=Rushy Pond,Rushy Pond      , 7
Up Type= 0
Dn Type= 0
Boundary for River Rch & Prof#=Rushy Pond,Rushy Pond      , 8
Up Type= 0
Dn Type= 0
Boundary for River Rch & Prof#=Wigwam Brook,Wigwam Brook    , 1
Up Type= 3
Up Slope=2.93038E-03
Dn Type= 0
Boundary for River Rch & Prof#=Wigwam Brook,Wigwam Brook    , 2
Up Type= 3
Up Slope=2.93038E-03
Dn Type= 0
Boundary for River Rch & Prof#=Wigwam Brook,Wigwam Brook    , 3
Up Type= 3
Up Slope=2.93038E-03
Dn Type= 0
Boundary for River Rch & Prof#=Wigwam Brook,Wigwam Brook    , 4
Up Type= 3
Up Slope=2.93038E-03
Dn Type= 0
Boundary for River Rch & Prof#=Wigwam Brook,Wigwam Brook    , 5
Up Type= 3
Up Slope=2.93038E-03
Dn Type= 0
Boundary for River Rch & Prof#=Wigwam Brook,Wigwam Brook    , 6
Up Type= 3
Up Slope=2.93038E-03
Dn Type= 0
Boundary for River Rch & Prof#=Wigwam Brook,Wigwam Brook    , 7
Up Type= 3
Up Slope=2.93038E-03
Dn Type= 0
Boundary for River Rch & Prof#=Wigwam Brook,Wigwam Brook    , 8
Up Type= 3
Up Slope=2.93038E-03
Dn Type= 0
Gate Openings=Exploits River  ,CB to BF4       ,43.309  ,Gate #1                         ,
    3.66      17    3.66      17    3.66      17    3.66      17    3.66      17
    3.66      17    3.66      17    3.66      17
Gate Openings=Exploits River  ,CB to BF4       ,43.2577 ,Outside Gate                    ,
  3.9624       1  3.9624       1  3.9624       1  3.9624       1  3.9624       1
  3.9624       1  3.9624       1  3.9624       1
Gate Openings=Exploits River  ,CB to BF4       ,43.2577 ,Obermeyer                       ,
     1.5       1     1.5       1     1.5       1     1.5       1     1.5       1
     1.5       1     1.5       1     1.5       1
Gate Openings=Exploits River  ,CB to BF4       ,43.231  ,Inside Gate                     ,
  2.1336       1  2.1336       1  2.1336       1  2.1336       1  2.1336       1
  2.1336       1  2.1336       1  2.1336       1
Gate Openings=Exploits River  ,CB to BF4       ,43.231  ,RCC Fboards                     ,
      .9       1      .9       1      .9       1      .9       1      .9       1
      .9       1      .9       1      .9       1
Gate Openings=Exploits River  ,BF3 to BF2      ,23.7635 ,BF Gates                        ,
   4.328       9   4.328       9   4.328       9   4.328       9   4.328       9
   4.328       9   4.328       9   4.328       9
Gate Openings=Exploits River  ,BF3 to BF2      ,23.7635 ,BF Fboards                      ,
    1.22       1    1.22       1    1.22       1    1.22       1    1.22       1
    1.22       1    1.22       1    1.22       1
DSS Import StartDate=01jun2019
DSS Import StartTime=24:00
DSS Import EndDate=08jun2019
DSS Import EndTime=00:00
DSS Import GetInterval= 0
DSS Import Interval=1DAY
DSS Import GetPeak= 1
DSS Import FillOption= 1
TSRecord= 1
TSRecord Loc=B1              ,B1              ,0.9685
TSRecord DssFilename=dss
TSRecord DssPathname=//SUBSTR1TOLITREDIND/FLOW/01JUN2019/1HOUR/RUN:100YEAR_SPILL_OPEN/
TSRecord End
TSRecord= 2
TSRecord Loc=Badger Brk      ,Badger Brk      ,1.9217
TSRecord DssFilename=dss
TSRecord DssPathname=//BADGER1/FLOW/01JUN2019/1HOUR/RUN:100YEAR_SPILL_OPEN/
TSRecord End
TSRecord= 3
TSRecord Loc=BF1             ,BF1             ,1.2372
TSRecord DssFilename=dss
TSRecord DssPathname=//SUBSTREAM5TOEXPL/FLOW/01JUN2019/1HOUR/RUN:100YEAR_SPILL_OPEN/
TSRecord End
TSRecord= 4
TSRecord Loc=BF2             ,BF2             ,1.2490
TSRecord DssFilename=dss
TSRecord DssPathname=//SUBSTREAM4RURAL/FLOW/01JUN2019/1HOUR/RUN:100YEAR_SPILL_OPEN/
TSRecord End
TSRecord= 5
TSRecord Loc=BF2             ,BF2             ,0.3773
TSRecord DssFilename=dss
TSRecord DssPathname=//SUBSTREAM4URBAN/FLOW/01JUN2019/1HOUR/RUN:100YEAR_SPILL_OPEN/
TSRecord End
TSRecord= 6
TSRecord Loc=BF3             ,BF3             ,2.1832
TSRecord DssFilename=dss
TSRecord DssPathname=//SUBSTREAM3RURAL/FLOW/01JUN2019/1HOUR/RUN:100YEAR_SPILL_OPEN/
TSRecord End
TSRecord= 7
TSRecord Loc=BF3             ,BF3             ,0.8646
TSRecord DssFilename=dss
TSRecord DssPathname=//SUBSTREAM3URBAN/FLOW/01JUN2019/1HOUR/RUN:100YEAR_SPILL_OPEN/
TSRecord End
TSRecord= 8
TSRecord Loc=BF4             ,BF4             ,0.9422
TSRecord DssFilename=dss
TSRecord DssPathname=//SUBSTREAM2RURAL/FLOW/01JUN2019/1HOUR/RUN:100YEAR_SPILL_OPEN/
TSRecord End
TSRecord= 9
TSRecord Loc=BF4             ,BF4             ,0.8648
TSRecord DssFilename=dss
TSRecord DssPathname=//SUBSTREAM2URBAN/FLOW/01JUN2019/1HOUR/RUN:100YEAR_SPILL_OPEN/
TSRecord End
TSRecord= 10
TSRecord Loc=Corduroy Brk    ,Corduroy Brk    ,3.8918
TSRecord DssFilename=dss
TSRecord DssPathname=//SUBCORDBROOK5RURAL/FLOW/01JUN2019/1HOUR/RUN:100YEAR_SPILL_OPEN/
TSRecord End
TSRecord= 11
TSRecord Loc=Corduroy Brk    ,Corduroy Brk    ,3.3476
TSRecord DssFilename=dss
TSRecord DssPathname=//SUBCORDUROYBROOK4/FLOW/01JUN2019/1HOUR/RUN:100YEAR_SPILL_OPEN/
TSRecord End
TSRecord= 12
TSRecord Loc=Corduroy Brk    ,Corduroy Brk    ,1.8184
TSRecord DssFilename=dss
TSRecord DssPathname=//SUBCORDUROYBROOK3/FLOW/01JUN2019/1HOUR/RUN:100YEAR_SPILL_OPEN/
TSRecord End
TSRecord= 13
TSRecord Loc=Corduroy Brk    ,Corduroy Brk    ,1.2395
TSRecord DssFilename=dss
TSRecord DssPathname=//SUBCORD2TONEWGAUGE/FLOW/01JUN2019/1HOUR/RUN:100YEAR_SPILL_OPEN/
TSRecord End
TSRecord= 14
TSRecord Loc=Exploits River  ,Mill to LRI     ,127.9419
TSRecord DssFilename=dss
TSRecord DssPathname=//EXPLOITSRIVER24/FLOW/01JUN2019/1HOUR/RUN:100YEAR_SPILL_OPEN/
TSRecord End
TSRecord= 15
TSRecord Loc=Exploits River  ,Mill to LRI     ,98.9083
TSRecord DssFilename=dss
TSRecord DssPathname=//SUBEXPLMILLTONOEL/FLOW/01JUN2019/1HOUR/RUN:100YEAR_SPILL_OPEN/
TSRecord End
TSRecord= 16
TSRecord Loc=Exploits River  ,Mill to LRI     ,75.9221
TSRecord DssFilename=dss
TSRecord DssPathname=//SUBEXPLNOELTOBAD/FLOW/01JUN2019/1HOUR/RUN:100YEAR_SPILL_OPEN/
TSRecord End
TSRecord= 17
TSRecord Loc=Exploits River  ,Badger to Wigwam,53.6747
TSRecord DssFilename=dss
TSRecord DssPathname=//SUBEXPLBAGERTOCHAR/FLOW/01JUN2019/1HOUR/RUN:100YEAR_SPILL_OPEN/
TSRecord End
TSRecord= 18
TSRecord Loc=Exploits River  ,Badger to Wigwam,51.6126
TSRecord DssFilename=dss
TSRecord DssPathname=//SUBSANDYBRKDAMTOEXPL/FLOW/01JUN2019/1HOUR/RUN:100YEAR_SPILL_OPEN/
TSRecord End
TSRecord= 19
TSRecord Loc=Exploits River  ,Badger to Wigwam,50.7343
TSRecord DssFilename=dss
TSRecord DssPathname=//SANDYBROOK1/FLOW/01JUN2019/1HOUR/RUN:100YEAR_SPILL_OPEN/
TSRecord End
TSRecord= 20
TSRecord Loc=Exploits River  ,RP to CB        ,46.8401
TSRecord DssFilename=dss
TSRecord DssPathname=//SUBEXPLCHARTOGOOD/FLOW/01JUN2019/1HOUR/RUN:100YEAR_SPILL_OPEN/
TSRecord End
TSRecord= 21
TSRecord Loc=Exploits River  ,CB to BF4       ,43.2587
TSRecord DssFilename=dss
TSRecord DssPathname=//SUBEXPLGOODTOGRAND/FLOW/01JUN2019/1HOUR/RUN:100YEAR_SPILL_OPEN/
TSRecord End
TSRecord= 22
TSRecord Loc=Exploits River  ,CB to BF4       ,41.6238
TSRecord DssFilename=dss
TSRecord DssPathname=//SUBEXPLGRFALLSTOST/FLOW/01JUN2019/1HOUR/RUN:100YEAR_SPILL_OPEN/
TSRecord End
TSRecord= 23
TSRecord Loc=Exploits River  ,CB to BF4       ,33.2970
TSRecord DssFilename=dss
TSRecord DssPathname=//SUBEXPLSTONYTOGRRATT/FLOW/01JUN2019/1HOUR/RUN:100YEAR_SPILL_OPEN/
TSRecord End
TSRecord= 24
TSRecord Loc=Exploits River  ,CB to BF4       ,31.6595
TSRecord DssFilename=dss
TSRecord DssPathname=//GREATRATTLINGBROOK1/FLOW/01JUN2019/1HOUR/RUN:100YEAR_SPILL_OPEN/
TSRecord End
TSRecord= 25
TSRecord Loc=Exploits River  ,CB to BF4       ,30.6038
TSRecord DssFilename=dss
TSRecord DssPathname=//SUBGRRATTTOEXPL/FLOW/01JUN2019/1HOUR/RUN:100YEAR_SPILL_OPEN/
TSRecord End
TSRecord= 26
TSRecord Loc=Exploits River  ,BF3 to BF2      ,23.7697
TSRecord DssFilename=dss
TSRecord DssPathname=//SUBEXPLGRRATTTOBISH/FLOW/01JUN2019/1HOUR/RUN:100YEAR_SPILL_OPEN/
TSRecord End
TSRecord= 27
TSRecord Loc=Exploits River  ,BF2 to BF1      ,21.7690
TSRecord DssFilename=dss
TSRecord DssPathname=//SUBEXPLBISHTOGAUGE/FLOW/01JUN2019/1HOUR/RUN:100YEAR_SPILL_OPEN/
TSRecord End
TSRecord= 28
TSRecord Loc=Exploits River  ,BF1 to Outlet   ,18.0852
TSRecord DssFilename=dss
TSRecord DssPathname=//SUBJUMPERSBROOK/FLOW/01JUN2019/1HOUR/RUN:100YEAR_SPILL_OPEN/
TSRecord End
TSRecord= 29
TSRecord Loc=Exploits River  ,BF1 to Outlet   ,9.3990
TSRecord DssFilename=dss
TSRecord DssPathname=//SUBEXPLNEWGAUTOOUT/FLOW/01JUN2019/1HOUR/RUN:100YEAR_SPILL_OPEN/
TSRecord End
TSRecord= 30
TSRecord Loc=Exploits River  ,BF1 to Outlet   ,8.4354
TSRecord DssFilename=dss
TSRecord DssPathname=//SUBEASTERN/FLOW/01JUN2019/1HOUR/RUN:100YEAR_SPILL_OPEN/
TSRecord End
TSRecord= 31
TSRecord Loc=Exploits River  ,BF1 to Outlet   ,3.1711
TSRecord DssFilename=dss
TSRecord DssPathname=//SUBOUTLET1/FLOW/01JUN2019/1HOUR/RUN:100YEAR_SPILL_OPEN/
TSRecord End
TSRecord= 32
TSRecord Loc=Exploits River  ,BF1 to Outlet   ,0.0989
TSRecord DssFilename=dss
TSRecord DssPathname=//SUBOUTLET2/FLOW/01JUN2019/1HOUR/RUN:100YEAR_SPILL_OPEN/
TSRecord End
TSRecord= 33
TSRecord Loc=GF1             ,GF1             ,4.002117
TSRecord DssFilename=dss
TSRecord DssPathname=//SUBPETERS4/FLOW/01JUN2019/1HOUR/RUN:100YEAR_SPILL_OPEN/
TSRecord End
TSRecord= 34
TSRecord Loc=GF1             ,GF1             ,3.1868
TSRecord DssFilename=dss
TSRecord DssPathname=//SUBPETERS3/FLOW/01JUN2019/1HOUR/RUN:100YEAR_SPILL_OPEN/
TSRecord End
TSRecord= 35
TSRecord Loc=GF1             ,GF1             ,1.3701
TSRecord DssFilename=dss
TSRecord DssPathname=//SUBPETERS2/FLOW/01JUN2019/1HOUR/RUN:100YEAR_SPILL_OPEN/
TSRecord End
TSRecord= 36
TSRecord Loc=GF1             ,GF1             ,0.0107
TSRecord DssFilename=dss
TSRecord DssPathname=//SUBPETERSRIV1TOOUTL/FLOW/01JUN2019/1HOUR/RUN:100YEAR_SPILL_OPEN/
TSRecord End
TSRecord= 37
TSRecord Loc=Little Red Ind  ,LRI to B1       ,1.4448
TSRecord DssFilename=dss
TSRecord DssPathname=//SUBLITTLEREDINDIAN/FLOW/01JUN2019/1HOUR/RUN:100YEAR_SPILL_OPEN/
TSRecord End
TSRecord= 38
TSRecord Loc=Little Rushy Pd ,Little Rushy Pd ,0.5608
TSRecord DssFilename=dss
TSRecord DssPathname=//SUBLITTLERUSHYPOND/FLOW/01JUN2019/1HOUR/RUN:100YEAR_SPILL_OPEN/
TSRecord End
TSRecord= 39
TSRecord Loc=Mullens Pond    ,Mullens Pond    ,0.4097
TSRecord DssFilename=dss
TSRecord DssPathname=//SUBSTREAM6TOSEWER/FLOW/01JUN2019/1HOUR/RUN:100YEAR_SPILL_OPEN/
TSRecord End
TSRecord= 40
TSRecord Loc=Rushy Pond      ,Rushy Pond      ,1.605
TSRecord DssFilename=dss
TSRecord DssPathname=//SUBTORUSHYATTCHBR/FLOW/01JUN2019/1HOUR/RUN:100YEAR_SPILL_OPEN/
TSRecord End
TSRecord= 41
TSRecord Loc=Wigwam Brook    ,Wigwam Brook    ,4.6443
TSRecord DssFilename=dss
TSRecord DssPathname=//SUBTOWIGWAMBRKCUL3/FLOW/01JUN2019/1HOUR/RUN:100YEAR_SPILL_OPEN/
TSRecord End
TSRecord= 42
TSRecord Loc=Wigwam Brook    ,Wigwam Brook    ,4.0688
TSRecord DssFilename=dss
TSRecord DssPathname=//SUBWIGWAMBRKCUL1TO3/FLOW/01JUN2019/1HOUR/RUN:100YEAR_SPILL_OPEN/
TSRecord End
DSS File=C:\Users\neuf58278\Desktop\Exploits\HECRAS\FloodMappingModel_temp\FloodMapModel\100Year_Spill_Open.dss
Storage Area Elev=Power Canal     , 8
   60.95      61   61.05   61.07  60.706  60.706  60.706  60.706
Storage Area Elev=Rushy Pond      , 8
      71      71      71      71      71      71      71      71
