HEC-RAS study Exploits_FMM.prj: Exploits_FMM

--- Exploits_FMM.g01 (geometry) --- (continued)

Type RM Length L Ch R = 6 ,3.1355  ,,,
BEGIN DESCRIPTION:
Earle Ave Lateral Structure
END DESCRIPTION:
Node Name=Overland Flood L
Lateral Weir Pos= 3
Lateral Weir Distance=170
Lateral Weir TW Multiple XS=0
Lateral Weir WD=2
Lateral Weir Coef=1.4
LW OverFlow Method 2D=0
LW OverFlow Use Velocity Into 2D=0
Lateral Weir WSCriteria=-1
Lateral Weir Flap Gates= 0
Lateral Weir Hagers EQN= 0 ,,,,,
Lateral Weir SS=0.05,0.05,
Lateral Weir Type= 0
Lateral Weir Connection Pos and Dist= 3 ,
Lateral Weir SE= 30
       0  83.488   4.792  83.252   8.626  81.932  18.578  82.657  68.911  82.319
  70.906  82.655 104.662  81.573 120.044  82.222 140.164  81.757 146.879  82.151
 154.352  81.755 168.593  82.679  177.35  82.416 184.189  81.612 192.047  81.637
 198.914  82.223 204.788  81.786 233.494  82.449  252.12  81.967  255.83  82.383
 261.752  81.527  266.59  81.443 271.195  82.185 275.183  81.914 279.857  82.566
 284.314  82.014 291.074  82.848 294.838   82.02 300.457  82.691  317.69  82.659
Lateral Weir Centerline= 6
     598784.0014     5423064.672     598785.8363     5423032.498
     598783.8728     5422967.001     598778.1891     5422934.955
     598725.5215     5422815.929         598704.        5422763.
LW Div RC= 0 ,False,,

Type RM Length L Ch R = 1 ,3.1255  ,140.89,141.34,141.87
BEGIN DESCRIPTION:
CB65 (SEM 2019)
END DESCRIPTION:
XS GIS Cut Line= 6
  599266.8888036 5422774.8046831  598968.7684036 5422985.7969831
  598947.8764036 5422996.1072831  598925.3868036 5423003.0525831
  598846.0789036 5423077.0938831  598785.5560036 5423054.6643831
#Sta/Elev= 30
       0   87.39  103.78   85.45  118.75   85.45  131.72   86.26   141.7   84.18
  151.68   83.75  202.57   83.62  226.52   84.13  268.43   83.57  291.39   84.42
  319.33   84.35  345.27   83.41  359.24   83.55  362.24   83.33  369.11   81.28
  396.13   80.39  401.86   78.72  403.13   79.77  406.37   80.57  411.08   81.29
  480.75   80.92  484.73   81.76  488.71   80.95  508.62   80.96  517.58   82.52
  526.52   81.34  533.47   81.87  539.43   81.07  565.25   82.08  585.11    81.9
#Mann= 3 , 0 , 0
       0     .06       0  396.13     .04       0  406.37     .06       0
Bank Sta=396.13,406.37
XS Rating Curve= 0 ,0
Exp/Cntr=0.3,0.1

Type RM Length L Ch R = 1 ,2.9841  ,132.18,130.08,127.31
BEGIN DESCRIPTION:
CB64 (SEM 2019)
END DESCRIPTION:
XS GIS Cut Line= 6
  599087.3422036 5422751.6271831  598880.7607036 5422892.9679831
  598841.3814036 5422913.4247831  598819.2225036 5422924.0081831
  598788.9800036 5422939.1293831  598781.0770036 5422946.2952831
#Sta/Elev= 30
       0   86.97   24.93   86.26   31.91   84.18    34.9   84.51   38.89   84.37
   41.88   83.47   44.88   83.15   67.81   83.32    73.8   82.86   81.77   82.87
   87.76    82.1   98.73   82.24  112.69   83.15  153.57   82.96  175.51   83.35
  226.37    81.8  237.34   82.39  244.32   81.49  249.31   81.38  290.74   81.26
  300.73   80.24  304.19   79.31   308.1   79.14  312.04   80.22  313.55   79.97
  321.23   81.28  341.12    81.6  355.05   81.24  360.81   82.21  363.72   82.06
#Mann= 3 , 0 , 0
       0     .06       0  300.73     .04       0  312.04     .06       0
Bank Sta=300.73,312.04
XS Rating Curve= 0 ,0
Exp/Cntr=0.3,0.1

Type RM Length L Ch R = 1 ,2.8540  ,57.31,59.87,61.24
BEGIN DESCRIPTION:
CB63 (SEM 2019)
END DESCRIPTION:
XS GIS Cut Line= 5
  599065.1171036 5422603.4601831  598784.4433036 5422788.5138831
  598776.8891036 5422798.9922831  598765.3136036 5422817.1823831
  598738.3420036 5422843.4443831
#Sta/Elev= 30
       0   87.95    6.98   88.03   16.96   86.41   28.93   85.73   69.83   85.43
  101.75   85.72  109.74   84.07  114.72   84.06  118.71   83.29  157.62   83.33
  228.45    82.4  239.42   82.95  286.31   83.56  321.23    83.3   332.2   82.72
  338.18   83.03  342.15   82.82   345.3   81.72  347.28   81.82  350.41   80.05
  353.33   78.82  354.49   79.14  355.83   78.69  359.65   79.75  362.16   80.31
  370.59   80.27  371.67    80.8  403.66   80.65  406.33   81.97  408.31   82.25
#Mann= 3 , 0 , 0
       0     .06       0  350.41     .04       0  359.65     .06       0
Bank Sta=350.41,359.65
XS Rating Curve= 0 ,0
Exp/Cntr=0.3,0.1

Type RM Length L Ch R = 1 ,2.7942  ,15.15,15.84,16.54
BEGIN DESCRIPTION:
CB62 (SEM 2019)
END DESCRIPTION:
XS GIS Cut Line= 4
  599037.6004036 5422570.6517831  598755.1677036 5422755.0008831
  598728.9333036 5422773.8567831  598714.1960036 5422786.4449831
#Sta/Elev= 30
       0   88.18    7.98   88.29   13.97   87.87   18.96   86.39   34.92   85.86
   42.91   86.13    47.9   85.49   98.79   85.55  102.78   85.31  106.77   84.48
  128.72    83.6   187.6   83.42  208.55   82.96  213.54   82.31  228.51   82.28
  242.48   83.01  285.38   83.43  319.31   83.44   325.3   83.06  331.29   83.97
  334.28   83.98  344.13   83.12  351.96   81.75   368.6   81.07  373.16   80.19
  377.76   79.01  382.63    79.3   384.6   80.29  386.57   81.91  388.96   82.01
#Mann= 3 , 0 , 0
       0     .06       0  373.16     .04       0   384.6     .06       0
Bank Sta=373.16,384.6
XS Rating Curve= 0 ,0
Exp/Cntr=0.3,0.1

Type RM Length L Ch R = 1 ,2.7783  ,193.4,194.01,193.92
BEGIN DESCRIPTION:
US of Harris Ave Culvert - CB61 (SEM 2019)
END DESCRIPTION:
XS GIS Cut Line= 4
  599003.7337036 5422521.9683831  598742.5944036 5422736.8439831
  598723.3109036 5422760.2968831  598707.1600036 5422771.1619831
#Sta/Elev= 30
       0   88.41   12.97   88.36   16.96   86.86   18.95   86.56   30.92    86.8
    40.9   86.49   70.83   84.72  116.72   84.24  145.65   83.29  208.49   83.08
  217.47   82.16  235.43   82.02  240.42   82.18   245.4   83.01  268.35   83.35
  321.22   83.01   331.2   83.73  339.16   82.47  347.97    82.7  354.83   82.07
  369.54   82.61  369.92   81.91  372.83   81.84  373.79   81.23  374.82   80.18
  377.64   79.26  381.08   79.83  383.76   81.26  385.52   82.16  388.01   82.67
#Mann= 3 , 0 , 0
       0     .06       0  373.79     .04       0  383.76     .06       0
Bank Sta=373.79,383.76
XS Rating Curve= 0 ,0
Exp/Cntr=0.3,0.1

Type RM Length L Ch R = 2 ,2.675   ,,,
Node Photo=.\Photos\CB-CR-12.JPG
BEGIN DESCRIPTION:
Harris Ave Culvert
END DESCRIPTION:
Node Name=CB-CR-12
Bridge Culvert--1,0,-1,-1, 0
Deck Dist Width WeirC Skew NumUp NumDn MinLoCord MaxHiCord MaxSubmerge Is_Ogee
6.5,185,1.4,0, 400, 400, , , 0.98, 0, 3,3,,
       0    .996   5.979   7.972   9.965  12.954  17.936  19.929  21.922  25.908
  29.894   30.89  35.873  37.866  42.848   47.83   50.82  54.805  59.788  63.774
  66.763  69.752  72.742   78.72  82.706  90.678   95.66  99.646 101.639 106.621
 108.614 109.611 111.604 114.593 116.586 119.575 122.565 124.558 128.544 133.485
 141.292 143.244 149.099 151.051 153.003  155.93 156.906  159.89 166.852 167.846
 172.819 173.813 175.802 179.781  181.77 182.764 184.753 190.721 193.704 197.682
 198.677 201.661 205.639 210.612 213.595 215.565 222.461 224.431 227.386 231.327
 236.252 238.222 241.177 244.133 245.118 253.983 256.939 265.834 266.826 267.818
 273.772 280.719 282.704 286.673 288.658 296.597 298.581 301.517 307.348 309.291
  314.15 316.094 318.038 319.981 321.925 322.897 326.784 327.755 329.699 331.641
 335.521 337.461 340.371 342.311 345.221 348.131 349.101 351.041 353.951 354.927
 355.902 356.877 358.827 359.802 361.752 363.702 364.678 366.628 368.578 370.524
 371.497 372.471 374.417  375.39 376.363 378.328 382.256 384.147 385.092 386.037
 388.873 390.849 392.825 394.801 396.767 401.658 402.636 406.549 408.506 410.462
 412.419 414.375 415.353  417.31 418.288 421.223 422.201 423.179 426.114 431.983
 432.961 434.918 436.874 438.831  441.45  444.25 445.214  447.14 449.067 450.031
 451.021 453.994 454.985 457.957 459.939  461.92 465.883 470.837 471.828 472.819
  473.81 475.791 476.782 477.773 480.745 481.736  486.69 488.672 491.644 493.626
 495.607 496.598 500.561 504.525 505.515 507.497 509.479  511.46 514.433 517.377
 518.354 520.307 521.284  522.26 526.167 527.144  528.12 530.074  531.05 533.004
 534.957  536.91  539.84 543.788 545.782  546.78 548.774 550.768  553.76 554.757
 556.751 559.743  560.74 562.734 564.729 566.723 568.717 570.712 571.709 573.703
 575.697 577.692 579.686 580.683 584.672 585.653 588.595 589.576 591.537 593.499
  595.46 596.441 599.383 601.345 602.326 605.268 607.229 609.191 610.172 612.133
 614.095 615.076 618.999 620.981 623.954 626.927 627.919 629.901 631.883 633.865
 635.847 637.829 639.812 641.794 643.776 645.758 646.749 648.731 650.714 652.695
 654.675 661.607 666.558 667.548 671.509  677.45 683.391 686.362 690.328 693.317
 695.309 696.305 699.293 700.289 703.278 707.262 711.247 712.243 714.235 716.227
 718.219 720.212 721.208   723.2 725.192 727.184 728.147 731.036 732.962 734.888
 736.814 739.703 741.628 743.554 746.443 751.258 753.203 755.168 758.115  760.08
  764.01 764.992 766.957  767.94 770.887 772.852 775.799 777.764  778.73 782.597
 784.531 785.498 787.431 789.365 791.298 793.231 794.198 796.132 799.032 801.932
 804.833 807.735 811.603 814.505 818.373 824.176  826.11  828.06 830.025 833.956
 836.904 837.886 839.852   842.8 844.765  847.74 850.715 852.699 855.674 857.658
 861.625 865.553 868.414 869.368 870.321 872.228 873.182 876.043 878.903 881.764
 882.718 884.713  885.71 888.702 890.697 892.692 895.684 897.679 901.669 904.661
 906.656 911.643 914.636 921.618 925.608 930.595 933.587 937.577 940.569 944.559
 952.539 955.531 958.523 960.518 961.515 962.513 964.508 966.503   967.5 969.495
 971.488 974.476 992.4011006.3421013.3131016.2931030.1831034.1521036.1361041.097
1046.0571048.042 1052.011054.9871056.9711064.9081070.8611076.8141078.7981083.759
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     -50 -49.004 -44.021 -42.028 -40.035 -37.046 -32.064 -30.071 -28.078 -24.092
 -20.106  -19.11 -14.127 -12.134  -7.152   -2.17     .82   4.805   9.788  13.774
  16.763  19.752  22.742   28.72  32.706  40.678   45.66  49.646  51.639  56.621
  58.614  59.611  61.604  64.593  66.586  69.575  72.565  74.558  78.544  83.485
  91.292  93.244  99.099 101.051 103.003  105.93 106.906  109.89 116.852 117.846
 122.819 123.813 125.802 129.781  131.77 132.764 134.753 140.721 143.704 147.682
 148.677 151.661 155.639 160.612 163.595 165.565 172.461 174.431 177.386 181.327
 186.252 188.222 191.177 194.133 195.118 203.983 206.939 215.834 216.826 217.818
 223.772 230.719 232.704 236.673 238.658 246.597 248.581 251.517 257.348 259.291
  264.15 266.094 268.038 269.981 271.925 272.897 276.784 277.755 279.699 281.641
 285.521 287.461 290.371 292.311 295.221 298.131 299.101 301.041 303.951 304.927
 305.902 306.877 308.827 309.802 311.752 313.702 314.678 316.628 318.578 320.524
 321.497 322.471 324.417  325.39 326.363 328.328 332.256 334.147 335.092 336.037
 338.873 340.849 342.825 344.801 346.767 351.658 352.636 356.549 358.506 360.462
 362.419 364.375 365.353  367.31 368.288 371.223 372.201 373.179 376.114 381.983
 382.961 384.918 386.874 388.831  391.45  394.25 395.214  397.14 399.067 400.031
 401.021 403.994 404.985 407.957 409.939  411.92 415.883 420.837 421.828 422.819
  423.81 425.791 426.782 427.773 430.745 431.736  436.69 438.672 441.644 443.626
 445.607 446.598 450.561 454.525 455.515 457.497 459.479  461.46 464.433 467.377
 468.354 470.307 471.284  472.26 476.167 477.144  478.12 480.074  481.05 483.004
 484.957  486.91  489.84 493.788 495.782  496.78 498.774 500.768  503.76 504.757
 506.751 509.743  510.74 512.734 514.729 516.723 518.717 520.712 521.709 523.703
 525.697 527.692 529.686 530.683 534.672 535.653 538.595 539.576 541.537 543.499
  545.46 546.441 549.383 551.345 552.326 555.268 557.229 559.191 560.172 562.133
 564.095 565.076 568.999 570.981 573.954 576.927 577.919 579.901 581.883 583.865
 585.847 587.829 589.812 591.794 593.776 595.758 596.749 598.731 600.714 602.695
 604.675 611.607 616.558 617.548 621.509  627.45 633.391 636.362 640.328 643.317
 645.309 646.305 649.293 650.289 653.278 657.262 661.247 662.243 664.235 666.227
 668.219 670.212 671.208   673.2 675.192 677.184 678.147 681.036 682.962 684.888
 686.814 689.703 691.628 693.554 696.443 701.258 703.203 705.168 708.115  710.08
  714.01 714.992 716.957  717.94 720.887 722.852 725.799 727.764  728.73 732.597
 734.531 735.498 737.431 739.365 741.298 743.231 744.198 746.132 749.032 751.932
 754.833 757.735 761.603 764.505 768.373 774.176  776.11  778.06 780.025 783.956
 786.904 787.886 789.852   792.8 794.765  797.74 800.715 802.699 805.674 807.658
 811.625 815.553 818.414 819.368 820.321 822.228 823.182 826.043 828.903 831.764
 832.718 834.713  835.71 838.702 840.697 842.692 845.684 847.679 851.669 854.661
 856.656 861.643 864.636 871.618 875.608 880.595 883.587 887.577 890.569 894.559
 902.539 905.531 908.523 910.518 911.515 912.513 914.508 916.503   917.5 919.495
 921.488 924.476 942.401 956.342 963.313 966.293 980.183 984.152 986.136 991.097
 996.057 998.042 1002.011004.9871006.9711014.9081020.8611026.8141028.7981033.759
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BR Coef=-1 , 0 , 0 ,, 0 ,,,0.8,-1,,0,
WSPro=,,,, 1 ,,,, 0 ,,,, 0 ,,,,-1 ,-1 ,-1 , 0 , 0 , 0 , 0 , 0
Culvert=1,1.8,,193,0.024,0.5,1,2,1,79.291,378,79.084,336,Culvert #1  , 0 ,1
     378     336
BC Culvert Barrel=1,1,0
Culvert Bottom n=0.024
BC Design=,, 0 ,, 0 ,,,,,,
BC Use User HTab Curves=0
BC User HTab FreeFlow(D)= 0

Type RM Length L Ch R = 1 ,2.5843  ,8.39,7.31,6.47
BEGIN DESCRIPTION:
DS of Harris Ave Culvert - CB55 (SEM 2019)
END DESCRIPTION:
XS GIS Cut Line= 6
  598912.7168036 5422404.4931831  598684.5476036 5422553.9206831
  598640.2977036 5422586.3329831  598623.7612036 5422596.5856831
  598592.2485036 5422616.1576831  598536.5895036 5422697.6742831
#Sta/Elev= 30
       0   88.58       5   88.45   15.99   87.13   38.96   85.16   42.96   85.32
   47.96   84.09   50.95   84.35  120.89   84.55  149.86   83.96  161.85   83.38
  182.83   82.91  297.68   81.67   325.6    82.2  331.18   81.82  333.29   80.67
   334.7   79.06  337.04   79.02  339.81   79.61  339.99   80.48  340.56   80.52
  342.18   81.48     350   82.04  355.88   81.55  374.52   81.28   399.3   81.67
   405.3   80.84  421.27   81.67  426.27   82.43  460.22   82.16  482.85   82.53
#Mann= 3 , 0 , 0
       0     .06       0  331.18     .04       0  342.18     .06       0
Bank Sta=331.18,342.18
XS Rating Curve= 0 ,0
Exp/Cntr=0.3,0.1

Type RM Length L Ch R = 1 ,2.5770  ,42.36,42.41,42.21
BEGIN DESCRIPTION:
CB54 (SEM 2019)
END DESCRIPTION:
XS GIS Cut Line= 6
  598879.9084036 5422374.8597831  598678.0383036 5422542.6368831
  598635.3367036 5422577.7340831  598620.1232036 5422593.2783831
  598591.6191036 5422611.8452831  598530.3116036 5422688.6821831
#Sta/Elev= 30
       0   88.78    6.99   88.39   31.94   85.94   41.92   84.27   68.87   84.08
   98.81   84.49  136.73   84.49  161.69   83.41  180.65   82.94  291.11   81.68
  316.78   82.17  324.13   81.68  324.95   81.26   327.5   79.34  329.51   79.21
   330.7   79.39     333   81.14  333.74   81.48  339.45   81.64  340.49   82.06
  347.29   82.16  350.21   81.72  359.92    81.4  389.52   81.76  394.51   80.82
   413.5   81.82   415.5   82.28  419.49   82.43  445.47   82.08  471.83   82.37
#Mann= 3 , 0 , 0
       0     .06       0  324.95     .04       0     333     .06       0
Bank Sta=324.95,333
XS Rating Curve= 0 ,0
Exp/Cntr=0.3,0.1

Type RM Length L Ch R = 1 ,2.5346  ,32.49,32.18,32.57
BEGIN DESCRIPTION:
CB53 (SEM 2019)
END DESCRIPTION:
XS GIS Cut Line= 6
  598840.4193036 5422350.5179831  598631.0253036 5422522.1264831
  598605.5711036 5422547.3068831  598592.6726036 5422560.8667831
  598578.0785036 5422602.4461831  598517.2877036 5422674.8868831
#Sta/Elev= 30
       0   88.17       4   87.88    7.99    88.2   19.98   86.12   24.98   85.79
   28.97   85.04  126.87   84.06   198.8   82.75  277.69   81.78  302.56   82.36
  311.78   81.76   312.6    81.4  314.52   79.44     316   78.85  317.35   79.17
  320.51   81.46  331.13   81.76  354.63    81.4  362.46   81.69  366.38   81.39
  374.31   81.92   383.3   81.86   385.3   81.75   387.3   80.95   389.3   80.76
  397.29   81.84  402.28   81.99  433.25   82.32  437.25   81.94  463.88   82.17
#Mann= 3 , 0 , 0
       0     .06       0   312.6     .04       0  320.51     .06       0
Bank Sta=312.6,320.51
XS Rating Curve= 0 ,0
Exp/Cntr=0.3,0.1

Type RM Length L Ch R = 1 ,2.5024  ,14.1,14.23,14.22
BEGIN DESCRIPTION:
CB52 (SEM 2019)
END DESCRIPTION:
XS GIS Cut Line= 6
  598823.8167036 5422327.2346831  598585.9026036 5422524.3086831
  598573.8210036 5422535.7313831  598566.2142036 5422543.6688831
  598510.3601036 5422593.7239831  598488.4919036 5422618.3471831
#Sta/Elev= 30
       0   90.01       2   89.57       7   87.61      11   86.89   24.99   86.45
   27.99   86.81   31.99   88.11   43.99    87.9   47.99   87.42   53.99   85.56
   58.99   84.95  106.98   83.68  150.97   83.83  259.95   82.91  286.94   82.14
  303.94    82.4  316.76   82.07  325.56   80.65  326.49   80.89  328.77   79.47
  330.71   78.64  332.36   78.87  332.53   79.25  333.03    79.4  335.71      81
  337.54   81.32  356.29   80.85  360.24   80.44  367.15   80.94  444.49   81.99
#Mann= 3 , 0 , 0
       0     .06       0  328.77     .04       0  333.03     .06       0
Bank Sta=328.77,333.03
XS Rating Curve= 0 ,0
Exp/Cntr=0.3,0.1

Type RM Length L Ch R = 1 ,2.4882  ,135.22,136.59,137.12
BEGIN DESCRIPTION:
US of Cromer Avenue Culvert - CB51 (SEM 2019)
END DESCRIPTION:
XS GIS Cut Line= 6
  598816.4083036 5422301.8345831  598577.3856036 5422508.3330831
  598561.2533036 5422529.4474831  598549.6777036 5422542.0151831
  598503.4702036 5422581.7887831  598485.4116036 5422601.9763831
#Sta/Elev= 30
       0   91.16       3   90.26       8      88      11   87.45   15.99   87.78
   26.99   87.74   30.99   87.19   40.98   87.01   72.97   87.07   79.97   87.38
   85.96   87.01   93.96   87.11   98.96   86.43  101.96   85.36  104.96    84.8
  109.95   84.17  147.94   84.29  289.88   82.91  341.46   81.54  343.79   80.56
  347.21   79.95  347.69   78.77  348.95   78.54  351.67    78.7  356.82   80.09
  361.53   80.63  370.52    80.9  421.49   81.58  432.48    82.1  447.58   81.99
#Mann= 3 , 0 , 0
       0     .06       0  347.21     .04       0  356.82     .06       0
Bank Sta=347.21,356.82
XS Rating Curve= 0 ,0
Exp/Cntr=0.3,0.1

Type RM Length L Ch R = 2 ,2.41    ,,,
Node Photo=.\Photos\CB-CR-11.JPG
BEGIN DESCRIPTION:
Cromer Avenue Culvert
END DESCRIPTION:
Node Name=CB-CR-11
Bridge Culvert--1,0,-1,-1, 0
Deck Dist Width WeirC Skew NumUp NumDn MinLoCord MaxHiCord MaxSubmerge Is_Ogee
4,128,1.4,0, 400, 400, , , 0.98, 0, 3,3,,
     111112.9864114.9728122.9184123.9116 125.898127.8844129.8708132.8504134.8368
136.8232139.8027142.7823145.7619147.7483149.7347153.7075155.6939158.6735160.6599
165.6259170.5919173.5817174.5783175.5749177.5682178.5648184.5444 185.541187.5343
190.5241194.5105196.5037198.4969199.4936201.4868204.4766 208.463209.4597211.4529
214.4427215.4393217.4325218.4291 221.419225.4054 226.402229.3918232.3716233.3633
238.3213240.3045243.2793245.2625247.2457250.2205251.2121254.1869257.1618259.1491
261.1406266.1194275.0813279.0643284.0431290.0177292.0092295.9922297.9837299.9753
301.9403303.8788305.8174308.7252 311.633314.5408316.4794321.3257323.2643325.2028
329.0799331.0185334.9821340.9275342.9093348.8547351.8274353.8092358.7637361.7364
362.7273   365.7366.6909368.6727369.6636371.6085375.4983377.4432 381.333385.2228
387.1677389.1126390.0851  392.03393.0024394.9692398.9462399.9405 401.929404.9118
407.8945409.8831412.8658415.8486417.8372418.8314421.8142424.7787429.6589430.6349
 432.587434.5391436.4911438.4432439.4193441.3713442.3474443.3234445.2755447.2275
449.1796450.1556451.1317453.0837456.9879458.9399 459.916462.8441463.8371466.8161
 470.788 473.767 477.739 479.725 482.704 485.683 486.676 489.655 491.641 493.627
494.6199496.6059500.5779505.5429510.5079511.5009515.4729517.4589518.4569520.4529
 521.451 522.449 524.445526.4411528.4371529.4352531.4312534.4253535.4233537.4193
539.4154540.4134542.4095543.4075544.4055545.3839547.3406550.2757553.2108554.1891
556.1458557.1242558.1026560.0593562.9944563.9727564.9511566.9078567.8862569.8429
573.7563577.6698581.6408583.6263 584.619587.5973594.5465595.5392598.5175599.5102
601.4957605.4667609.4377612.4159615.3942618.3724621.3506622.3434623.3362627.3071
630.2854633.2717634.2672 636.258639.2443643.2261646.2124647.2078649.1987650.1942
651.1896654.1759655.1713658.1576663.1348664.1302666.1211670.1028672.0938673.0892
675.0801678.0663679.0618682.0481 684.039692.9979694.9888 699.966701.9568704.9432
705.9386 706.934708.9167712.8821714.8647722.7954724.7781726.7607728.7434730.7261
732.7087734.6915737.6655738.6568739.6481740.6395741.6308743.6135745.5961746.5875
748.5701750.5528751.5441754.5182755.5095759.4749762.4489763.4402765.4229768.3969
770.3795773.3535776.3276777.3189779.3016783.2669785.2496786.2409788.2236790.2062
791.1976794.1794 800.174803.1714804.1705807.1678 809.166812.1634815.1607816.1599
819.1572821.1554825.1519826.1509  827.15830.1474832.1456833.1447835.1429843.1359
845.1341847.1323850.1296852.1279854.1261855.1252857.1234858.1225861.1199863.1181
865.1163872.0981873.0913881.0366885.0092888.9819891.9613892.9545894.9408897.9203
899.9066904.8773907.8715909.8676910.8657911.8638913.8599 915.856919.8483922.8425
924.8386927.8328 930.827934.8193937.8135938.8115941.8057943.8019944.7999947.7941
948.7922951.7864953.7825955.7786959.7709 961.767963.7632964.7612966.7574968.7535
970.7496  975.74977.7361980.7303985.7206989.7129990.7109995.7013997.6974999.6935
 1001.691002.6881004.6841007.6781013.6661014.6651015.6631017.6591022.6491023.647
1026.6411030.634 1032.631034.626 1037.621039.6161041.6121044.6061046.6031047.601
1049.5971052.5911054.5871058.5791061.5741064.5681069.5581071.5541072.5521074.548
1078.5411080.5371082.5331086.525 1089.521090.5171092.5141093.512 1094.511101.496
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     193194.9864196.9728204.9184205.9116 207.898209.8844211.8708214.8504216.8368
218.8232221.8027224.7823227.7619229.7483231.7347235.7075237.6939240.6735242.6599
247.6259252.5919255.5817256.5783 257.575259.5681260.5648266.5444 267.541269.5342
272.5241276.5105278.5037280.4969281.4936283.4868286.4766 290.463291.4597293.4529
296.4427297.4393299.4325300.4291 303.419307.4054 308.402311.3918314.3716315.3633
320.3213322.3045325.2793327.2625329.2457332.2205333.2121336.1869339.1618341.1491
343.1406348.1194357.0813361.0643366.0431372.0177374.0092377.9922379.9837381.9753
383.9403385.8788387.8174390.7252 393.633396.5408398.4794403.3257405.2643407.2028
411.0799413.0185416.9821422.9275424.9093430.8547433.8274435.8092440.7637443.7364
444.7273   447.7448.6909450.6727451.6636453.6085457.4983459.4432 463.333467.2228
469.1677471.1126472.0851  474.03475.0024476.9692480.9462481.9405 483.929486.9118
489.8945491.8831494.8658497.8486499.8372500.8314503.8142506.7787511.6589512.6349
 514.587516.5391518.4911520.4432521.4193523.3713524.3474525.3234527.2755529.2275
531.1796532.1556533.1317535.0837538.9879540.9399 541.916544.8441545.8371548.8161
 552.788 555.767 559.739 561.725 564.704 567.683 568.676 571.655 573.641 575.627
576.6199578.6059582.5779587.5429592.5079593.5009597.4729599.4589600.4569602.4529
 603.451 604.449 606.445608.4411610.4371611.4352613.4312616.4253617.4233619.4193
621.4154622.4134624.4095625.4075626.4055627.3839629.3406632.2757635.2108636.1891
638.1458639.1242640.1026642.0593644.9944645.9727646.9511648.9078649.8862651.8429
655.7563659.6698663.6408665.6263 666.619669.5973676.5465677.5392680.5175681.5102
683.4957687.4667691.4377694.4159697.3942700.3724703.3506704.3434705.3362709.3071
712.2854715.2717716.2672 718.258721.2443725.2261728.2124729.2078731.1987732.1942
733.1896736.1759737.1713740.1576745.1348746.1302748.1211752.1028754.0938755.0892
757.0801760.0663761.0618764.0481 766.039774.9979776.9888 781.966783.9568786.9432
787.9386 788.934790.9167794.8821796.8647804.7954806.7781808.7607810.7434812.7261
814.7087816.6915819.6655820.6568821.6481822.6395823.6308825.6135827.5961828.5875
830.5701832.5528833.5441836.5182837.5095841.4749844.4489845.4402847.4229850.3969
852.3795855.3535858.3276859.3189861.3016865.2669867.2496868.2409870.2236872.2062
873.1976876.1794 882.174885.1714886.1705889.1678 891.166894.1634897.1607898.1599
901.1572903.1554907.1519908.1509  909.15912.1474914.1456915.1447917.1429925.1359
927.1341929.1323932.1296934.1279936.1261937.1252939.1234940.1225943.1199945.1181
947.1163954.0981955.0913963.0366967.0092970.9819973.9613974.9545976.9408979.9203
981.9066986.8773989.8715991.8676992.8657993.8638995.8599 997.8561001.8481004.843
1006.8391009.8331012.8271016.8191019.8131020.8121023.8061025.802  1026.81029.794
1030.7921033.7861035.7821037.7791041.7711043.7671045.7631046.7611048.7571050.754
 1052.75 1057.741059.736 1062.731067.7211071.7131072.7111077.7011079.6971081.693
 1083.691084.6881086.6841089.6781095.6661096.6651097.6631099.6591104.6491105.647
1108.6411112.634 1114.631116.626 1119.621121.6161123.6121126.6061128.6031129.601
1131.5971134.5911136.5871140.5791143.5741146.5681151.5581153.5541154.5521156.548
1160.5411162.5371164.5331168.525 1171.521172.5171174.5141175.512 1176.511183.496
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BR Coef=-1 , 0 , 0 ,, 0 ,,,0.8,-1,,0,
WSPro=,,,, 1 ,,,, 0 ,,,, 0 ,,,,-1 ,-1 ,-1 , 0 , 0 , 0 , 0 , 0
Culvert=1,1.5,,134,0.024,0.9,1,2,3,78.431,349,77.839,432.5,Culvert #1  , 0 ,1
     349   432.5
BC Culvert Barrel=1,Barrel 1,0
Culvert Bottom n=0.024
BC Design=,, 0 ,, 0 ,,,,,,
BC Use User HTab Curves=0
BC User HTab FreeFlow(D)= 0

Type RM Length L Ch R = 1 ,2.3516  ,21.57,23.16,24.6
BEGIN DESCRIPTION:
DS of Cromer Avenue Culvert - CB47A (SEM 2019)
END DESCRIPTION:
XS GIS Cut Line= 6
  598814.8208036 5422283.3137831  598463.9485036 5422471.2181831
  598439.3462036 5422475.7369831  598428.4321036 5422480.3671831
  598396.7289036 5422512.8974831  598380.5929036 5422540.9687831
#Sta/Elev= 30
       0   90.09    7.98   89.91   13.97   88.33   32.92   88.25   42.89   87.04
   93.77   87.14   98.76   86.45   122.7      86  127.69   85.62  133.67   83.53
  184.55   84.83  213.47   84.94  290.28   83.76  315.22   83.09  318.22    82.2
   326.2   82.42  344.15   81.45  351.13   82.53  362.11   82.93   416.3   83.07
  423.03   82.52  424.02   82.18  424.61   81.13   432.3   77.93   441.8    79.9
  444.76   81.15  447.73   81.94  475.37   81.91  482.31    84.7  512.69   83.35
#Mann= 3 , 0 , 0
       0     .06       0  424.61     .04       0  444.76     .06       0
Bank Sta=424.61,444.76
XS Rating Curve= 0 ,0
Exp/Cntr=0.3,0.1

Type RM Length L Ch R = 1 ,2.3284  ,54.28,51.41,47.74
BEGIN DESCRIPTION:
CB47 (SEM 2019)
END DESCRIPTION:
XS GIS Cut Line= 6
  598806.8833036 5422270.0844831  598466.1847036 5422457.5424831
  598445.1671036 5422458.3405831  598430.6150036 5422457.0176831
  598403.7920036 5422461.4068831  598368.7474036 5422524.4549831
#Sta/Elev= 30
       0    89.6   29.99   88.58   33.99   87.43   91.97   87.16   96.97   86.32
  121.96   85.85  126.96   84.19  137.95   84.22  141.95   83.55  179.94   84.77
  246.91   84.66   303.9   83.29  309.89   82.12  361.88   81.14  373.87   82.88
  393.65   83.65  411.85   83.08  419.64   78.84  423.09    77.7  424.36   78.55
  434.22   78.35  441.98   83.23  449.75   82.87  458.68   85.02  463.67   82.33
  500.62   81.82  506.61    83.4  514.59   87.59  518.88   85.99  523.82   86.09
#Mann= 3 , 0 , 0
       0     .06       0  411.85     .04       0  441.98     .06       0
Bank Sta=411.85,441.98
XS Rating Curve= 0 ,0
Exp/Cntr=0.3,0.1

Type RM Length L Ch R = 1 ,2.2770  ,109.14,107.44,105.29
BEGIN DESCRIPTION:
CB46 (SEM 2019)
END DESCRIPTION:
XS GIS Cut Line= 6
  598748.6748036 5422228.8094831  598437.9404036 5422382.6762831
  598410.4405036 5422410.7154831  598403.1644036 5422420.3066831
  598385.6653036 5422445.4461831  598349.5527036 5422514.4237831
#Sta/Elev= 30
       0   87.86   50.96   87.04   58.96   85.86   89.93   86.11  106.92   84.94
  147.89   83.89  191.86   83.87  202.85   84.35  236.83   83.76  255.81   84.37
  281.79   83.85  309.77   84.15  316.77   83.05  323.76   82.92  329.76   82.11
  342.75   81.99  360.49   78.69  387.87   76.81  394.28   75.74  401.02   76.87
  405.96      77  413.87   82.57  419.79   83.14  443.68   80.84  481.66   80.49
  495.65   79.22  498.65   79.57  499.65   82.13  500.65   82.59  506.55   82.16
#Mann= 3 , 0 , 0
       0     .06       0  387.87     .04       0  401.02     .06       0
Bank Sta=387.87,401.02
XS Rating Curve= 0 ,0
Exp/Cntr=0.3,0.1

Type RM Length L Ch R = 1 ,2.1696  ,140.3,140.79,140.92
BEGIN DESCRIPTION:
CB45 (SEM 2019)
END DESCRIPTION:
XS GIS Cut Line= 4
598319.4898035985422302.89758309598304.6069035995422412.36908309
598304.6069035995422441.47338309598284.1017035985422472.23118309
#Sta/Elev= 30
       0   77.94   13.93   77.78   23.89   77.33   28.86   77.54   37.82   77.37
   39.81   77.59   59.72   76.99   70.67   77.03   80.62   76.73   82.61      77
   87.59   76.43   90.57   76.82  104.51   77.49  107.49   77.98  112.29   77.25
   113.5    77.3  114.59   76.76   117.1   76.28  118.27   75.89  124.17   75.63
  126.62   76.07     136   77.21  139.58   77.32  140.58   77.75  146.58   77.66
  151.57   78.45  153.57    79.5  156.57   80.41  158.57   80.64  176.55    80.4
#Mann= 3 , 0 , 0
       0     .12       0   117.1     .04       0  126.62     .12       0
Bank Sta=117.1,126.62
XS Rating Curve= 0 ,0
Exp/Cntr=0.3,0.1

Type RM Length L Ch R = 1 ,2.0288  ,109.29,107.77,103.25
BEGIN DESCRIPTION:
CB44 (SEM 2019)
END DESCRIPTION:
XS GIS Cut Line= 5
598267.9260035995422274.58248309598169.9077035985422412.66408309
598168.0155035985422436.18168309598166.3618035985422454.37178309
598165.3697035985422493.06718309
#Sta/Elev= 30
       0   77.81   90.64   76.81   96.62   76.96   99.61    78.1   101.6   77.85
  103.59   76.77  105.58   77.47  109.57   76.48  119.53   76.73  125.51   76.27
  133.48    77.3  143.44   75.41  159.37   76.61  163.36   78.36  165.35   78.62
   171.3   78.25   177.2   77.01  180.15    75.9  186.05    75.4  192.87   75.58
  200.52   74.71  202.88   74.99  204.06   75.74  205.39   75.79  208.33   77.37
  212.19   78.14   223.1   78.43  226.08   78.05  235.01   78.89   249.9    78.7
#Mann= 3 , 0 , 0
       0     .06       0  192.87     .04       0  204.06     .06       0
Bank Sta=192.87,204.06
XS Rating Curve= 0 ,0
Exp/Cntr=0.3,0.1

Type RM Length L Ch R = 1 ,1.9210  ,103.73,102.63,101.07
BEGIN DESCRIPTION:
CB43 (SEM 2019)
END DESCRIPTION:
XS GIS Cut Line= 6
598141.9840035985422175.89268309598071.0043035985422334.94178309
598089.3018035985422373.01228309598097.5700035985422384.91858309
598107.9798035985422442.61798309598146.2174035985422509.26838309
#Sta/Elev= 30
       0   77.45   10.95   77.45   15.92      77   22.89   77.59   29.86   76.93
    41.8   76.92   48.77   76.44   89.57   76.67   99.52   76.25  102.51   76.63
  108.48   76.05  173.17   76.58  217.37   76.12   217.7   75.69  220.16   75.49
  222.29   74.04  230.05    75.7   230.9   76.36  234.88   76.75  251.77   76.24
  282.58   76.47  286.55   77.36  288.54   76.69  294.52   76.74  298.52   77.34
   307.5   77.12  317.48   77.53   354.4   77.23  359.39   77.47  366.37   78.81
#Mann= 3 , 0 , 0
       0     .06       0   217.7     .04       0  230.05     .06       0
Bank Sta=217.7,230.05
XS Rating Curve= 0 ,0
Exp/Cntr=0.3,0.1

Type RM Length L Ch R = 1 ,1.8184  ,7.84,8.26,8.68
BEGIN DESCRIPTION:
CB42 (SEM 2019)
END DESCRIPTION:
XS GIS Cut Line= 6
598136.1632035985422177.48018309597998.8662035995422422.63288309
598011.5803035985422443.45768309598024.4788035985422452.38738309
598069.8827035995422481.36228309598140.9257035985422518.79338309
#Sta/Elev= 30
       0   77.38      24   77.36      31    76.8      53   76.34   87.99   76.62
   93.99   75.94  132.99   76.35  156.99   76.41  168.99   76.07  202.99   76.29
  230.98   75.86  232.98   75.03  238.98   74.15  239.98    74.2  242.98   75.28
  248.98   76.09  309.25   74.95  310.69      74  311.81    73.8   313.6   74.23
  314.69   74.97  321.07   75.59  334.04   76.08  345.01   75.74  352.99   76.27
  360.97   76.11  374.93    76.8   447.3   77.29  450.27   77.43  455.23   78.56
#Mann= 3 , 0 , 0
       0     .06       0  309.25     .04       0  314.69     .06       0
Bank Sta=309.25,314.69
XS Rating Curve= 0 ,0
Exp/Cntr=0.3,0.1

Type RM Length L Ch R = 1 ,1.8101  ,28.7,29.33,29.9
BEGIN DESCRIPTION:
US of Duggan Street 2 Culvert - CB41 (SEM 2019)
END DESCRIPTION:
XS GIS Cut Line= 6
598133.0940035985422178.43268309597992.2276035995422430.28798309
598004.9657035985422447.42648309598017.8642035985422459.00198309
598066.9365035985422486.87738309598141.9840035985422531.49338309
#Sta/Elev= 30
       0   77.33   27.96   77.17   31.95   76.59   42.94   76.38   81.88   76.34
   86.87   76.67   90.87   75.96   134.8   76.48  165.75   76.07   201.7    76.3
  227.66   75.85  235.65   74.15  238.65   74.44  242.64   75.74  245.64   76.13
  307.99   75.22  314.98   74.83  316.65   74.01  318.43   73.58  319.14   73.58
  321.63   74.89  327.26   75.35  361.91   76.22   372.8   76.01  399.57   76.58
  404.53   77.01  406.51   76.78  452.15   77.23  464.06   78.02     471   78.02
#Mann= 3 , 0 , 0
       0     .06       0  314.98     .04       0  321.63     .06       0
#XS Ineff= 2 , 0
             242    75.8
Permanent Ineff=
       T       F
Bank Sta=314.98,321.63
XS Rating Curve= 0 ,0
Exp/Cntr=0.3,0.1

Type RM Length L Ch R = 2 ,1.798   ,,,
Node Photo=.\Photos\CB-CR-10.JPG
BEGIN DESCRIPTION:
Duggan Street 2 Culvert
END DESCRIPTION:
Node Name=CB-CR-10
Bridge Culvert--1,0,-1,-1, 0
Deck Dist Width WeirC Skew NumUp NumDn MinLoCord MaxHiCord MaxSubmerge Is_Ogee
5,13,1.4,0, 400, 400, , , 0.98, 0, 3,3,,
     -87-85.0058-83.0116-81.0174-79.0232-78.0261-76.0319-75.0348-73.0406-72.0435
-69.0522 -67.058-64.0667-63.0696-61.0754-60.0783-56.0899-53.0986-51.1044-50.1073
-48.1131 -47.116-45.1218-44.1247-41.1334-40.1363-39.1392-37.1451-35.1509-33.1567
-31.1625-30.1654-28.1712-27.1741-24.1828-22.1886-21.1915-19.1973-18.2002-17.2031
 -16.206-14.2118-13.2147-12.2176-9.22636-8.22926-6.23506-4.24087-3.24377-2.24667
-1.24957 -.25247  .74463 2.73882 3.73592 4.73302 6.72721 8.72141 9.7185111.71271
 13.7069 15.7011 16.6982 18.6924 19.6895 20.6866 21.6837 22.6808 23.6745 24.6683
 25.6621 26.6558 28.6434 30.6309 32.6184 33.6122  34.606 36.5935 37.5873 41.5623
 45.5374 46.5311 48.5187 49.5124 52.4937 54.4813 56.4688 57.4626 58.4563 60.4439
 61.4376 62.4314 63.4252  68.394 71.3753  72.369 73.3628 74.3566 76.3441 79.3254
 81.3129 82.3067 83.3004 84.2942  85.288 86.2818 88.2693  89.263 90.2568 94.2319
 96.2194 99.2007100.1945105.1633109.1384111.1259112.1196114.1072115.1009116.0947
117.0885 119.076122.0573123.0511124.0448126.0323127.0261131.0012131.9949132.9887
136.9638137.9575138.9513139.9451141.9326144.9139145.9077148.8889150.8765153.8578
154.8515156.8391158.8266160.8223161.8201163.8157164.8136165.8114167.8071169.8027
171.7984174.7918175.7897176.7875177.7853178.7832 179.781180.7788182.7745184.7701
 185.768187.7636189.7593191.7549194.7484195.7462197.7419199.7376200.7354201.7332
 202.731203.7289204.7267206.7224207.7202 208.718211.7115212.7094213.7072 214.705
216.7007218.6963 220.692221.6898222.6876224.6833225.6811226.6789227.6768228.6746
229.6602230.6459231.6315232.6172233.6028234.5885235.5741236.5598237.5454238.5311
239.5167240.5023 241.488243.4593244.4449245.4306246.4162247.4019248.3875249.3732
250.3588251.3445252.3301253.3157254.3014 255.287256.2727257.2583 258.244259.2296
260.2153261.2009262.1866264.1579265.1435266.1292267.1148268.1004269.0861270.0717
 272.043273.0287274.0143     275275.9856276.9713277.9569278.9425279.9282 280.901
281.8737282.8465 284.792285.7648286.7375288.6831289.6559290.6286291.6014292.5741
293.5469295.4924296.4652 297.438299.3835300.3562 301.329302.3018303.2745305.2201
306.1928307.1916308.1903 309.189310.1877311.1864312.1852313.1839314.1826315.1813
316.1801317.1788318.1775319.1762 320.175321.1737322.1724323.1711324.1604325.1497
 326.139327.1283328.1176329.1069330.0963331.0855332.0749333.0641334.0535335.0428
 336.032337.0214338.0107339.9893340.9786341.9679342.9572344.9358345.9251347.9037
 348.893349.8823350.8622 351.842352.8218353.8017355.7614356.7412358.7009359.6807
360.6606361.6404362.6202363.6001364.5799365.5598366.5396367.5194368.4993369.4791
 370.459371.4388372.4186374.3783375.3582 376.338377.3178378.2977379.2775380.2574
381.2372 382.217383.1969384.1767388.0961390.0558391.0356392.0155392.9953394.9735
 395.972396.9704397.9688398.9672399.9656 400.964401.9624402.9608403.9592 405.956
406.9544408.9512409.9496413.9433415.9401416.9385417.9369418.9353419.9337421.9305
423.9273424.9257426.9225428.9194429.9178430.9161 432.913433.9114434.9098435.9082
436.9066438.9034440.9002441.8986 442.897445.8923446.8906  447.89448.8892450.8878
 451.887453.8856455.8842457.8828460.8806461.8798463.8784464.8777466.8762468.8748
469.8741470.8734472.8719473.8712474.8705477.8683479.8669480.8661481.8654482.8647
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       0   1.994   3.988   5.983   7.977   8.974  10.968  11.965  13.959  14.956
  17.948  19.942  22.933   23.93  25.925  26.922   30.91  33.901  35.896  36.893
  38.887  39.884  41.878  42.875  45.867  46.864  47.861  49.855  51.849  53.843
  55.837  56.835  58.829  59.826  62.817  64.811  65.808  67.803    68.8  69.797
  70.794  72.788  73.785  74.782  77.774  78.771  80.765  82.759  83.756  84.753
   85.75  86.748  87.745  89.739  90.736  91.733  93.727  95.721  96.719  98.713
 100.707 102.701 103.698 105.692  106.69 107.687 108.684 109.681 110.675 111.668
 112.662 113.656 115.643 117.631 119.618 120.612 121.606 123.594 124.587 128.562
 132.537 133.531 135.519 136.512 139.494 141.481 143.469 144.463 145.456 147.444
 148.438 149.431 150.425 155.394 158.375 159.369 160.363 161.357 163.344 166.325
 168.313 169.307   170.3 171.294 172.288 173.282 175.269 176.263 177.257 181.232
 183.219 186.201 187.195 192.163 196.138 198.126  199.12 201.107 202.101 203.095
 204.089 206.076 209.057 210.051 211.045 213.032 214.026 218.001 218.995 219.989
 223.964 224.958 225.951 226.945 228.933 231.914 232.908 235.889 237.877 240.858
 241.852 243.839 245.827 247.822  248.82 250.816 251.814 252.811 254.807 256.803
 258.798 261.792  262.79 263.788 264.785 265.783 266.781 267.779 269.775  271.77
 272.768 274.764 276.759 278.755 281.748 282.746 284.742 286.738 287.735 288.733
 289.731 290.729 291.727 293.722  294.72 295.718 298.712 299.709 300.707 301.705
 303.701 305.696 307.692  308.69 309.688 311.683 312.681 313.679 314.677 315.675
  316.66 317.646 318.632 319.617 320.603 321.589 322.574  323.56 324.545 325.531
 326.517 327.502 328.488 330.459 331.445 332.431 333.416 334.402 335.388 336.373
 337.359 338.345  339.33 340.316 341.301 342.287 343.273 344.258 345.244  346.23
 347.215 348.201 349.187 351.158 352.144 353.129 354.115   355.1 356.086 357.072
 359.043 360.029 361.014     362 362.986 363.971 364.957 365.943 366.928 367.901
 368.874 369.847 371.792 372.765 373.738 375.683 376.656 377.629 378.601 379.574
 380.547 382.492 383.465 384.438 386.384 387.356 388.329 389.302 390.275  392.22
 393.193 394.192  395.19 396.189 397.188 398.186 399.185 400.184 401.183 402.181
  403.18 404.179 405.178 406.176 407.175 408.174 409.172 410.171  411.16  412.15
 413.139 414.128 415.118 416.107 417.096 418.086 419.075 420.064 421.054 422.043
 423.032 424.021 425.011 426.989 427.979 428.968 429.957 431.936 432.925 434.904
 435.893 436.882 437.862 438.842 439.822 440.802 442.761 443.741 445.701 446.681
 447.661  448.64  449.62   450.6  451.58  452.56  453.54 454.519 455.499 456.479
 457.459 458.439 459.419 461.378 462.358 463.338 464.318 465.298 466.278 467.257
 468.237 469.217 470.197 471.177 475.096 477.056 478.036 479.016 479.995 481.974
 482.972  483.97 484.969 485.967 486.966 487.964 488.962 489.961 490.959 492.956
 493.954 495.951  496.95 500.943  502.94 503.939 504.937 505.935 506.934 508.931
 510.927 511.926 513.923 515.919 516.918 517.916 519.913 520.911  521.91 522.908
 523.907 525.903   527.9 528.899 529.897 532.892 533.891  534.89 535.889 537.888
 538.887 540.886 542.884 544.883 547.881  548.88 550.878 551.878 553.876 555.875
 556.874 557.873 559.872 560.871 561.871 564.868 566.867 567.866 568.865 569.865
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BR Coef=-1 , 0 , 0 ,, 0 ,,,0.8,-1,,0,
WSPro=,,,, 1 ,,,, 0 ,,,, 0 ,,,,-1 ,-1 ,-1 , 0 , 0 , 0 , 0 , 0
Culvert=1,1.8,,23.8,0.024,0,1,2,3,73.775,318.5,73.569,405,Culvert #1  , 0 ,1.5
   318.5     405
BC Culvert Barrel=1,Barrel 1,0
Culvert Bottom n=0.024
BC Design=,, 0 ,, 0 ,,,,,,
BC Use User HTab Curves=0
BC User HTab FreeFlow(D)= 0

Type RM Length L Ch R = 1 ,1.7808  ,4,4.12,4.1
BEGIN DESCRIPTION:
DS of Duggan Street 2 Culvert - CB40 (SEM 2019)
END DESCRIPTION:
XS GIS Cut Line= 6
  598127.2732036 5422181.8722831  597931.0840036 5422325.8893831
  597952.3565036 5422389.3101831  597987.7173036 5422431.2258831
  597991.0750036 5422474.2155831  598128.0669036 5422562.3438831
#Sta/Elev= 30
       0   77.24  272.33   74.99  300.28   74.89  384.96   75.56   396.8   75.25
  399.68   74.72  400.39   74.83  401.46   74.66  403.15   73.78  404.89   73.65
  406.42   73.71   407.6   74.68  408.55   74.78   434.2   75.04  442.12   74.28
  447.07   74.18  458.96   75.36  468.86    75.6  471.83   75.18  482.75   75.58
  490.73   75.52  498.72   76.12  509.69   76.11  518.68   76.72  535.64   76.81
  547.62   76.43   556.6    76.9  568.58    77.1  572.57   77.94  576.56   78.08
#Mann= 3 , 0 , 0
       0     .06       0  400.39     .04       0  408.55     .06       0
Bank Sta=400.39,408.55
XS Rating Curve= 0 ,0
Exp/Cntr=0.3,0.1

Type RM Length L Ch R = 1 ,1.7767  ,36.56,39.97,45.4
BEGIN DESCRIPTION:
CB39 (SEM 2019)
END DESCRIPTION:
XS GIS Cut Line= 6
  598120.9232036 5422182.9305831  597928.0678036 5422324.6193831
  597978.8380036 5422465.2858831  598108.6602036 5422559.2667831
  598177.8398036 5422648.3882831  598042.4330036 5422887.5253831
#Sta/Elev= 30
       0   77.16  270.11      75  375.72   75.59  390.14   75.25  394.97   74.54
  401.22   73.58  403.37   74.01  409.02   73.85  410.52   74.47  455.83   75.33
   481.5    75.2  511.38   75.97  519.34   76.63  567.14   77.05  573.39      78
  581.38   78.28  615.32   78.31  620.32   79.69  675.23   79.81  713.21   79.23
   718.2   79.61   727.2   79.39  733.19   78.35  859.11   77.42   867.1   77.97
  890.09   78.16  897.08   78.78  904.08   80.35  921.07   82.39  945.05   84.01
#Mann= 3 , 0 , 0
       0     .06       0  394.97     .04       0  410.52     .06       0
Bank Sta=394.97,410.52
XS Rating Curve= 0 ,0
Exp/Cntr=0.3,0.1

Type RM Length L Ch R = 1 ,1.7367  ,72.93,74.53,73.28
BEGIN DESCRIPTION:
CB38 (SEM 2019)
END DESCRIPTION:
XS GIS Cut Line= 6
  598113.5148036 5422184.5180831  597925.0515036 5422323.0318831
  597944.4190036 5422391.6913831  597977.5650036 5422434.0527831
  597854.0535036 5422588.4321831  597761.0024036 5422804.3840831
#Sta/Elev= 30
       0   77.13  263.61   75.04  368.82   75.73  376.62   75.09  378.68   74.97
  384.97   72.75  387.06   73.07   387.3   73.82  390.89   73.84  393.04   74.44
  403.04   74.14  428.03    74.7  436.02   74.25  439.02   74.75  463.01   74.57
  475.01   75.06  478.01   74.69  534.98   75.79  542.98   76.72  547.97   76.36
  552.97   77.19  556.97   76.73  561.28   77.82  575.23   78.18   583.2   79.54
  628.04   80.27  641.99   81.42  676.86   82.29  700.78   83.83  793.44   88.03
#Mann= 3 , 0 , 0
       0     .06       0  376.62     .04       0  393.04     .12       0
Bank Sta=376.62,393.04
XS Rating Curve= 0 ,0
Exp/Cntr=0.3,0.1

Type RM Length L Ch R = 1 ,1.6622  ,89.74,90.38,91.64
BEGIN DESCRIPTION:
CB37 (SEM 2019)
END DESCRIPTION:
XS GIS Cut Line= 6
  598094.1470036 5422195.4495831  597921.8765036 5422322.0793831
  597938.5288036 5422376.2708831  597926.8710036 5422388.9844831
  597905.0853036 5422407.4081831  597793.3683036 5422542.7646831
#Sta/Elev= 30
       0   76.85   72.93   76.22   103.9   76.34  276.25   74.86  280.08   75.04
  283.91   74.85  287.75   74.16  300.75   73.85  302.64   73.34  304.88   73.46
  307.14   72.62  307.76   72.75  308.67   73.47  312.37   73.24  313.27   73.64
  315.16   73.32   316.3   73.96  336.28   74.39  347.27   73.99  349.27   74.42
  371.24   74.62  380.23   74.36   390.2   74.96  393.19   74.61  402.15   75.06
  423.07   74.59  446.98   74.71  472.88   76.64  483.84   78.63  491.81    78.4
#Mann= 3 , 0 , 0
       0     .06       0  300.75     .04       0   316.3     .12       0
Bank Sta=300.75,316.3
XS Rating Curve= 0 ,0
Exp/Cntr=0.3,0.1

Type RM Length L Ch R = 1 ,1.5718  ,7.97,8.23,8.18
BEGIN DESCRIPTION:
CB36 (SEM 2019)
END DESCRIPTION:
XS GIS Cut Line= 6
598130.9774035985422153.82638309597912.7666035985422314.15108309
597892.1868035985422320.75698309597875.9811035985422326.37938309
597762.7183035985422352.44538309597695.4723035985422424.76028309
#Sta/Elev= 30
       0   77.64       4   77.74    7.99   77.16  109.91   76.44  161.87   75.74
  288.46   75.38  289.86    74.9  293.72   74.41  296.47   73.26  299.99   73.22
  301.11   72.85  302.67   71.81  303.77   71.88  305.11   73.01  313.52   73.95
  318.49   73.74  328.42   74.36  332.39   73.75  335.37   74.42  339.35   74.61
  343.32   74.02  404.91   74.43  410.87   73.82   421.8   74.15  432.75   75.67
  441.73   75.82  444.72   76.17  450.71   78.42   453.7   79.04  524.52   80.04
#Mann= 3 , 0 , 0
       0     .06       0  299.99     .04       0  305.11     .12       0
Bank Sta=299.99,305.11
XS Rating Curve= 0 ,0
Exp/Cntr=0.3,0.1

Type RM Length L Ch R = 1 ,1.5636  ,5.61,5.41,5.26
BEGIN DESCRIPTION:
US of Duggan Street 1 Bridge - CB35 (SEM 2019)
END DESCRIPTION:
XS GIS Cut Line= 6
598134.6815035995422146.41808309597907.2213035985422308.62528309
597888.2181035985422314.14238309597873.0045035985422318.77258309
597758.8748035985422345.49718309597694.4140035995422411.53108309
#Sta/Elev= 30
       0   78.04   10.98   77.77   13.97   77.18  112.75   76.56  163.63    75.8
  250.44   75.42  260.42   75.07  284.32   75.44  299.16   75.06  303.99   73.39
  305.42   72.66  307.51   72.54  308.13   72.19  308.66   72.96  309.82   73.27
  312.66   73.08  316.06    74.1  319.04   74.35     324   73.87  334.93   73.72
  348.84   74.27  405.46   74.34  412.41    73.8  426.32   74.66  432.28   75.68
  452.13   76.13  454.11   76.59  458.08   78.68  460.06   79.22  524.56   79.78
#Mann= 3 , 0 , 0
       0     .06       0  303.99     .04       0  309.82     .12       0
Bank Sta=303.99,309.82
XS Rating Curve= 0 ,0
Exp/Cntr=0.3,0.1
