HEC-RAS study Exploits_FMM.prj: Exploits_FMM

--- Exploits_FMM.g01 (geometry) --- (continued)

Type RM Length L Ch R = 1 ,51.6126 ,1028.2,878.28,1098.98
BEGIN DESCRIPTION:
Sandy Brook - R01A (SEM 2019)
END DESCRIPTION:
XS GIS Cut Line= 6
  591015.8073036 5421847.6606831  590961.2592036 5421802.1725831
  590603.6302036 5421128.4707831  590615.2180036 5421046.1969831
  590961.0350036 5419812.3059831  590916.9701036 5419367.6498831
#Sta/Elev= 30
     -68   72.76  -50.24   69.19  -22.62   71.11   32.96   69.18  215.73   71.54
   321.6   71.61  355.56   69.22  519.35   72.14   796.7   70.91  801.82   67.69
  811.66   67.16  853.13   69.46 1079.99   70.55 1094.08   66.87 1131.62   66.38
 1385.35   67.42 1409.79   70.34 1659.55   70.11 1768.01   67.48 1813.39   70.54
 1914.14   69.37 1981.97   69.37 2083.72   69.86  2116.8   67.18 2136.61   71.24
 2142.61   73.63 2297.55    77.7 2512.48   93.26 2552.46   93.59 2577.45   90.82
#Mann= 10 ,-1 , 0
     -68     .12       0   796.7     .04       0  853.13     .12       0
 1079.99     .04       0 1409.79     .12       0 1659.55     .04       0
 1813.39     .12       0 1914.14     .04       0 1981.97     .12       0
 2136.61     .12       0
Bank Sta=796.7,2136.61
XS Rating Curve= 0 ,0
Exp/Cntr=0.3,0.1

Type RM Length L Ch R = 1 ,50.7343 ,828.8,921.88,912.98
BEGIN DESCRIPTION:
R02 (RIS 2013)
END DESCRIPTION:
XS GIS Cut Line= 4
  591299.4412036 5421388.9714831  591301.4423036 5421358.0241831
  591524.8619036 5420941.5243831  591978.0932036 5419658.0781831
#Sta/Elev= 30
     -27    71.5   49.94   70.87  209.75   73.34  247.71    70.6   256.7   70.54
  260.69   72.16  375.13   70.46  389.54   70.46  395.53   69.25  396.33   67.14
  405.56  65.168  425.06  66.458  535.38  67.178  788.35  67.208  846.47  65.878
  967.73  66.828  984.76  65.848 1051.08  67.088 1124.36  65.898 1141.96  67.908
    1152   70.82 1166.08   71.17 1258.93    73.5 1360.87    71.8  1468.8   72.08
 1555.74   77.56 1718.64   78.26  1769.6   81.82  1772.6   80.68 1837.56   82.62
#Mann= 3 , 0 , 0
     -27     .12       0  375.13     .04       0 1166.08     .12       0
Bank Sta=375.13,1166.08
XS Rating Curve= 0 ,0
Exp/Cntr=0.3,0.1

River Reach=Exploits River  ,Wigwam to RP
Reach XY= 30
     592433.2195      5420942.03      592470.065    5420951.3545
     592482.2928    5420954.4551     592517.7109    5420963.4103
     592550.0097    5420971.5845     592554.2749    5420972.6705
     592609.5446    5420986.6564     592675.4122     5420981.714
     592704.3074    5420979.5546     592753.5405     5420975.863
     592754.7815    5420975.7694     592755.2421    5420975.7254
     592758.2646    5420975.5052     592772.2769    5420974.4498
     592807.9881    5420971.7801     592809.8398    5420971.6345
     592812.8423    5420971.4141     592834.6414    5420969.7812
     592922.0496    5420923.5869     592967.1283    5420899.7529
      592985.806    5420889.8898     592992.7134    5420886.2312
     592993.5893    5420885.7728     593054.4258    5420853.6171
     593215.7868     5420692.619     593228.2796    5420680.1448
     593234.1458    5420674.3026     593251.6742    5420656.8053
     593300.4695     5420608.123593328.5783616975420580.42338077

Type RM Length L Ch R = 1 ,49.8124 ,803.52,523.74,378.79
BEGIN DESCRIPTION:
R02A (SEM 2019)
END DESCRIPTION:
XS GIS Cut Line= 4
592295.5420035985422017.53628309592416.5131035985421462.56678309
592540.6005035985420663.98338309592643.2720035995419696.13978309
#Sta/Elev= 30
       0   75.59  118.79   72.57  313.45   72.86  328.42   70.97  373.34   72.72
  387.32   71.03  450.21   76.44  473.17   74.49   512.1   74.77  528.07   70.01
  568.53   69.43  865.61   67.24  949.41   65.04 1024.24   66.55 1030.53   69.23
 1039.52   70.78 1090.46   70.53 1094.46   69.28  1139.1   65.94 1244.66   67.65
 1299.48    66.2 1310.23   69.95 1357.62   70.73  1447.1   73.33 1488.07   72.09
 1883.77   73.41 1996.69   78.37 2161.56   78.78 2286.47   82.17 2349.43   85.62
#Mann= 5 ,-1 , 0
       0     .12       0  568.53     .04       0 1030.53     .12       0
 1094.46     .04       0 1357.62     .12       0
Bank Sta=568.53,1357.62
XS Rating Curve= 0 ,0
Exp/Cntr=0.3,0.1

Type RM Length L Ch R = 1 ,49.2887 ,782.52,939.38,745.21
BEGIN DESCRIPTION:
Camp Island - R02A (SEM 2019)
END DESCRIPTION:
XS GIS Cut Line= 4
592978.1684035985421615.36878309593198.8770035985421269.38198309
592870.4438035985420655.51768309592904.3578035985420008.33668309
#Sta/Elev= 30
       0   74.77   94.86   73.45  100.85   71.71  104.84   73.24  124.81   73.64
  140.79   76.89  178.73   73.87  183.73   75.15  239.64   75.78  246.63   75.11
  252.62   72.12  426.39   69.61  521.26    69.3 535.519  63.705  553.78  66.665
 582.291  66.985 610.158  65.435 749.501  67.175 819.419  64.945 961.121  66.465
  993.69   67.11 1021.16   70.79 1122.57   73.34 1285.33   71.02 1379.19   72.36
 1615.84   77.92  1647.8   82.16 1677.75   83.77 1725.68   84.14 1754.64    81.6
#Mann= 3 , 0 , 0
       0     .12       0  426.39     .04       0 1021.16     .12       0
Bank Sta=426.39,1021.16
XS Rating Curve= 0 ,0
Exp/Cntr=0.3,0.1

River Reach=Exploits River  ,RP to CB
Reach XY= 30
593328.5783616975420580.42338077     593771.6442    5420128.9175
     593902.7783     5420059.881     594021.5076    5420044.5053
      594148.221    5420065.2206     594320.5165    5420160.6177
     594521.8948    5420296.6032      594775.297    5420500.9961
     594867.7145    5420555.1266      594958.337    5420583.8262
     595021.9304     5420576.204     595130.3235    5420541.6444
     595200.9614    5420481.2007     595258.9587     5420416.351
     595368.9978    5420417.7991      595484.828    5420461.6589
     595564.5394    5420515.6122     595660.6287    5420612.1266
     595910.7423    5420905.3672      596040.209    5421038.2871
     596364.6602    5421311.3488       596513.46    5421423.3657
     596719.2446    5421546.7115     596903.2042    5421559.7117
     596990.1651    5421546.0378     597169.0854    5421459.5021
      597233.264    5421407.4423     597308.4932    5421319.5417
     597369.1672    5421212.4015597386.2387024965421161.31664681

Type RM Length L Ch R = 1 ,48.3493 ,323.78,401.12,495.42
BEGIN DESCRIPTION:
Grand Falls Golf Club - R03 (RIS 2013)
END DESCRIPTION:
XS GIS Cut Line= 4
594097.2124035985420723.51688309593722.7239035985420282.07668309
593591.9733035985420171.52808309593462.8692035985420037.68388309
#Sta/Elev= 30
       0   79.53  271.95   78.03  354.93   72.73  491.91   71.43   520.9   72.44
   531.9   70.84   540.9    71.5  555.89   69.41  566.73   69.97  580.88   70.58
  583.87   69.29  585.64  66.995  586.71  68.465  595.59  66.225   600.6  69.065
  601.87  63.705  603.84  68.045  610.67  65.565  619.81  65.275  629.63  62.985
  648.77  64.935     695  64.605   734.6  65.985  750.26  67.815  750.39    71.6
  759.11   78.75  763.11   79.51  855.09   79.86  892.09   81.48  936.08   79.41
#Mann= 3 , 0 , 0
       0     .12       0  566.73     .04       0  750.39     .12       0
Bank Sta=566.73,750.39
XS Rating Curve= 0 ,0
Exp/Cntr=0.3,0.1

Type RM Length L Ch R = 1 ,47.9482 ,466.43,519.18,595.07
BEGIN DESCRIPTION:
DS of Rushy Pond Brook - R04 (RIS 2013)
END DESCRIPTION:
XS GIS Cut Line= 4
594169.7219035985420692.43048309594013.3890035985420154.02098309
593979.8898035995419678.27508309594038.2769035995419422.95438309
#Sta/Elev= 30
       0   76.81  126.92   73.51  274.83   73.45  373.77   71.15   550.7   70.53
  556.65    70.7  585.14   66.41  679.43   65.11   709.3   63.52  742.57   65.76
  793.33   66.46  798.37   68.61  804.61   73.82  810.16    76.2  817.61   77.32
   841.6   77.35   894.6   75.16  916.59   73.15 1034.57    72.6 1060.56   73.67
 1069.56   76.75 1073.56    77.1 1081.56   77.25 1085.56   75.69 1097.55    76.2
  1227.5   85.86 1277.49   91.46 1283.48   93.84 1286.48   92.92 1299.48   94.48
#Mann= 3 , 0 , 0
       0     .12       0   550.7     .04       0  810.16     .12       0
Bank Sta=550.7,810.16
XS Rating Curve= 0 ,0
Exp/Cntr=0.3,0.1

Type RM Length L Ch R = 1 ,47.4290 ,648.13,613.51,432.68
BEGIN DESCRIPTION:
R04A (SEM 2019)
END DESCRIPTION:
XS GIS Cut Line= 4
  594429.2282036 5421129.4479831  594228.1445036 5420880.7390831
  594282.1953036 5420653.8590831  594720.9810036 5419724.6056831
#Sta/Elev= 30
       0    83.7   39.98   89.44  135.93   88.56   194.9   91.29  240.87   90.93
  387.61    83.7  408.54   81.52  427.47    76.7   450.4   73.98     726   72.77
  785.98   72.13  807.97   70.47  837.01  66.985  854.51  68.645  854.67  66.695
  857.35  65.365  857.78  67.875  865.58  68.575  917.32  64.685 1029.05  65.365
 1043.41  64.285 1084.79  65.445 1096.67  68.185 1119.86   70.37 1145.85   74.71
 1312.79   78.14 1534.71    89.7  1561.7   88.46  1565.7   90.03  1580.7   91.33
#Mann= 3 , 0 , 0
       0     .12       0  807.97     .04       0 1119.86     .12       0
Bank Sta=807.97,1119.86
XS Rating Curve= 0 ,0
Exp/Cntr=0.3,0.1

Type RM Length L Ch R = 1 ,46.8155 ,102.81,43,165.09
BEGIN DESCRIPTION:
R05 (RIS 2013)
END DESCRIPTION:
XS GIS Cut Line= 6
  595151.1957036 5420826.9782831  594966.0689036 5420742.0971831
  594997.5544036 5420671.7178831  594967.9210036 5420499.2091831
  594876.3750036 5420390.4651831  594835.6290036 5420202.8752831
#Sta/Elev= 30
       0   84.15  154.61   78.81  163.48   77.22  216.69   77.65  225.69   75.03
  229.31  68.377 257.622  68.377 279.346  65.187 287.609  66.059 291.251  62.497
 309.362  67.255 338.582  63.963 363.374  67.265 372.458  64.273 380.855  67.291
 389.559   62.13 522.952  68.688 581.808  63.592 593.717  66.448 640.569  68.896
  644.85   75.96  651.82   79.34  661.77   78.34  674.71      83  684.66   81.17
  693.62   82.99   697.6   80.96  722.48    81.4   780.2   85.95  798.12   83.52
#Mann= 3 , 0 , 0
       0     .12       0  229.31     .04       0 640.569     .12       0
Bank Sta=229.31,640.569
XS Rating Curve= 0 ,0
Exp/Cntr=0.3,0.1

Type RM Length L Ch R = 5 ,46.780  ,,,
Node Photo=.\Photos\Goodyears Dam.JPG
BEGIN DESCRIPTION:
Goodyear's Dam
END DESCRIPTION:
Node Name=GY Dam
IW Pilot Flow=0
#Inline Weir SE= 30
     228  70.795 230.859  70.789 231.631  69.864 255.648  69.864 256.089  70.546
 260.282  70.569 262.695  69.044 408.695  69.044 409.516  68.584 461.516  68.584
 461.616  69.165 464.473  69.371  472.09  70.985 496.617  72.013 499.562  72.503
 508.395  72.205 514.284   72.56 546.061  72.523 557.865  72.995 582.374   72.82
 585.356  73.173 594.301  73.227  617.13    74.7 651.793  78.175 660.725  79.607
 663.703  80.588 694.376  81.992 713.165   82.08 736.899  81.592 784.313  81.752
IW Dist,WD,Coef,Skew,MaxSub,Min_El,Is_Ogee,SpillHt,DesHd
16,3.65,2.5,0,0.98,, 0 ,,,3,3,
Inline Weir Flap Gates= 0
IW Outlet Rating Curve= 0 ,False,,

Type RM Length L Ch R = 1 ,46.7725 ,238.71,238.6,356.06
BEGIN DESCRIPTION:
DS of Goodyear's Dam
END DESCRIPTION:
XS GIS Cut Line= 4
  595176.4633036 5420836.8297831  595037.1861036 5420663.0153831
  594997.4579036 5420440.5965831  594891.0985036 5420230.1995831
#Sta/Elev= 30
       0   84.99   68.92   84.08   76.91   81.97   98.88   71.99  111.87   68.27
  190.12   68.81  203.75   71.12  222.73    66.3 257.326  65.422 263.582  63.963
 288.374  67.265 297.458  64.273 305.855  67.291 314.559   62.13 382.608  65.452
  399.68   67.49  403.68   66.58  413.12   70.47  437.67   70.21  453.67   71.59
  475.64   69.83  479.64    67.6  491.63   64.53   511.6   64.49  521.59   65.19
  532.58   69.82  549.57   71.19  560.55   74.53  605.51   80.76  684.42   80.81
#Mann= 3 , 0 , 0
       0     .12       0  190.12    .035       0  413.12     .12       0
Bank Sta=190.12,413.12
XS Rating Curve= 0 ,0
Exp/Cntr=0.3,0.1

Type RM Length L Ch R = 1 ,46.5339 ,317.86,423.87,565.51
XS GIS Cut Line= 6
  595274.0180036 5420823.7344831  595239.7875036 5420555.3472831
  595238.4646036 5420486.5554831  595212.3369036 5420440.5839831
  595201.4228036 5420411.8104831  595203.4965036 5420001.7937831
#Sta/Elev= 30
       0   85.96   55.98   83.23   79.97   74.39   96.97   69.08  104.97   67.78
  252.92   67.21  262.03   65.43  266.87    69.4  270.84   69.03  273.83   66.19
  275.83   65.68  289.79   64.73  347.63    64.4  352.62   65.63  376.56   64.36
  384.54   65.29  451.21   64.64  457.19   67.08  466.16   66.21  471.14   64.34
  475.13   65.46  478.12   64.38     515  61.902     545  61.902  590.49   65.12
  610.08   67.49     642   68.26  736.74   67.06  807.55   78.84  833.48   81.61
#Mann= 3 , 0 , 0
       0     .12       0  262.03    .035       0  590.49     .12       0
Bank Sta=262.03,590.49
XS Rating Curve= 0 ,0
Exp/Cntr=0.3,0.1

Type RM Length L Ch R = 1 ,46.1100 ,800.96,791.92,793.35
BEGIN DESCRIPTION:
R07 (RIS 2013)
END DESCRIPTION:
XS GIS Cut Line= 4
595453.4822035985420727.51768309595538.1372035985420606.40498309
595665.5410035985420454.63808309595776.1744035995420329.63758309
#Sta/Elev= 30
       0   82.07   17.97   80.98   30.95   80.96   36.94   80.01   45.93   79.67
   49.92    78.9   66.89   77.48   74.88   75.54   98.84   67.65  104.83   66.52
  137.67   66.08  142.77   66.24  147.77   64.73  150.75   63.33  162.68  61.982
  196.65  62.412  201.42  62.062  273.43  61.362  333.52  62.612  334.97   63.49
  340.75    65.3  344.92   66.31  355.92   67.48   381.9   67.89   401.9   69.63
  425.88   74.82  452.87   79.89  468.87   81.15  484.86   83.89  512.85    84.7
#Mann= 3 , 0 , 0
       0     .12       0  137.67    .035       0  340.75     .12       0
Bank Sta=137.67,340.75
XS Rating Curve= 0 ,0
Exp/Cntr=0.3,0.1

Type RM Length L Ch R = 1 ,45.3181 ,604.09,552.23,528.89
BEGIN DESCRIPTION:
R08 (RIS 2013)
END DESCRIPTION:
XS GIS Cut Line= 2
595842.4030035995421461.21828309596295.4702035985420927.48878309
#Sta/Elev= 30
       0    78.7   42.94   76.64    73.9   74.03  125.84   71.94  224.71   71.36
  251.68   72.21  266.66   71.27  283.63   67.32  314.91   64.59  322.58   64.25
  330.57   66.21  336.57   66.48  344.56   65.47  353.48  62.551  372.73  61.831
  373.75  61.081  378.92  60.211  380.22  60.761  390.49  59.991  473.45  61.551
     497  61.131   551.1  62.041  559.28   63.89   573.2   72.98  577.26   74.83
  580.25   75.35  594.23   74.95  628.19   78.49  691.11   80.11   700.1   79.24
#Mann= 3 , 0 , 0
       0     .12       0  314.91    .035       0   573.2     .12       0
Bank Sta=314.91,573.2
XS Rating Curve= 0 ,0
Exp/Cntr=0.3,0.1

Type RM Length L Ch R = 1 ,44.7659 ,541.81,410.11,274.04
BEGIN DESCRIPTION:
R09 (RIS 2013)
END DESCRIPTION:
XS GIS Cut Line= 4
596246.1248035985422054.90958309596516.1615035985421558.45688309
596622.0283035985421353.49208309596761.9062035985421218.82748309
#Sta/Elev= 30
       0   78.34   13.98   78.58   18.97   76.82  113.83    77.9  125.81   77.09
  136.79   78.87  158.76   78.73  164.75   76.84  173.74    78.3  280.57   77.07
   459.3   70.55  510.23   70.13   528.2   67.21  548.52   65.75  561.15   62.87
  596.29  60.462  654.83  61.002  682.13  59.702  756.92  61.492  765.13  63.022
  785.05  61.452  800.87   62.59  807.78   64.32  824.71   73.15  833.67    75.2
  925.28   76.85  939.22   78.02  963.12   83.72  976.06   84.25     990   82.89
#Mann= 3 , 0 , 0
       0     .06       0  548.52    .035       0  800.87     .12       0
Bank Sta=548.52,800.87
XS Rating Curve= 0 ,0
Exp/Cntr=0.3,0.1

Type RM Length L Ch R = 1 ,44.3558 ,524.36,400.64,344.37
BEGIN DESCRIPTION:
First Falls
END DESCRIPTION:
XS GIS Cut Line= 4
     597278.6605     5422194.348      597007.465     5421671.309
     596869.2199     5421371.006     596764.6875     5421205.026
#Sta/Elev= 30
       0   78.62   16.98   70.37   28.96   70.51   46.93   68.67   61.91   69.84
  151.79   69.21  161.77   68.72  169.76    66.1  179.75    65.2  313.56   64.22
  326.54   64.95  330.53   64.06  336.52   66.82  346.51   66.92   351.5    64.9
  358.49   64.16  483.32   63.92  506.28    65.2  531.25   63.69  578.18    64.1
  586.17   63.85  589.17   62.71  596.16   62.09  903.41   62.43  923.75   62.84
   934.7   66.87  971.54   70.79 1056.18   75.03 1102.97   80.95 1115.92   80.93
#Mann= 3 , 0 , 0
       0     .06       0  589.17    .035       0  903.41     .12       0
Bank Sta=589.17,903.41
XS Rating Curve= 0 ,0
Exp/Cntr=0.3,0.1

Type RM Length L Ch R = 1 ,43.9551 ,107.68,95.97,20.95
BEGIN DESCRIPTION:
R11 (RIS 2013)
END DESCRIPTION:
XS GIS Cut Line= 3
597687.3123035985421827.51058309597121.5261035985421148.34858309
597054.8230035985421150.64028309
#Sta/Elev= 30
       0   72.05  101.99   71.22  111.99   70.08  123.99   71.78  146.99   71.93
  203.99   67.16  218.99   67.27  253.99   64.61  277.98    64.8  285.98   63.48
  306.01   63.02  316.98   62.09  319.98   60.77  334.15  59.054  338.84  56.754
  342.79  56.614  351.16  57.764  371.89  57.904  647.13  57.894  669.64  58.794
  700.34  57.744  863.07  57.684  879.31  58.344  880.69  59.714  883.73  60.514
  884.95   64.23  905.87   70.77   924.8   74.46  935.75   79.06   950.7   81.79
#Mann= 3 , 0 , 0
       0     .06       0  306.01    .035       0  884.95     .12       0
Bank Sta=306.01,884.95
XS Rating Curve= 0 ,0
Exp/Cntr=0.3,0.1

Type RM Length L Ch R = 1 ,43.8591 ,10.55,63.54,29.49
BEGIN DESCRIPTION:
Grand Falls Headpond
END DESCRIPTION:
XS GIS Cut Line= 5
  597643.7841036 5421540.2596831  597552.7011036 5421537.6815831
  597565.6518036 5421412.1162831  597114.0350036 5421122.2995831
  597052.4352036 5421142.5266831
#Sta/Elev= 30
   -25.7   77.55    -4.9   76.69   27.78   68.48    46.6   64.84    57.5   64.47
   61.46    65.3   63.44   64.85   96.23   64.51  137.98   62.05  147.92   60.65
  184.69   60.68  281.73  56.585   287.6  56.665  293.06  57.855  353.48  57.275
  392.73  58.125  409.26  57.495  448.75  57.385  512.54  58.045  652.95  57.455
  683.07  57.845  697.08   60.71  703.18   60.91  707.18   64.12  712.17   66.29
  726.16   70.28  744.11   74.13   749.1   75.89  775.04   81.01  792.99   82.43
#Mann= 3 , 0 , 0
   -25.7     .06       0  147.92    .035       0  697.08     .12       0
Bank Sta=147.92,697.08
XS Rating Curve= 0 ,0
Exp/Cntr=0.3,0.1

Type RM Length L Ch R = 1 ,43.7956 ,316.97,138.53,124.09
BEGIN DESCRIPTION:
Grand Falls Headpond
END DESCRIPTION:
XS GIS Cut Line= 6
  597730.0174036 5421503.0686831  597556.6698036 5421532.5221831
  597580.1693036 5421382.0480831  597466.4252036 5421254.2706831
  597113.7601036 5421095.2694831  597047.5184036 5421134.6734831
#Sta/Elev= 30
  -135.5   80.27  -79.55   79.19   -34.6    77.1   14.36   66.0625.35001   64.43
   37.33   65.31   86.12   64.42  150.82   60.86  231.79   60.69  257.24  58.105
  312.72  57.505  330.66  56.485  339.89  57.785  392.14  57.015  428.12  58.285
  442.99  57.295  667.17  57.405  692.32  57.865  705.95  61.165  706.87   60.71
  711.42   60.87  715.41   63.93  725.39   67.89  733.37   68.78  752.31   73.13
  758.27   73.55  780.01   71.92  791.87   73.32  810.64   78.81  832.38   81.05
#Mann= 3 , 0 , 0
  -135.5     .06       0  150.82    .035       0  706.87     .12       0
Bank Sta=150.82,706.87
XS Rating Curve= 0 ,0
Exp/Cntr=0.3,0.1

River Reach=Exploits River  ,CB to BF4
Reach XY= 30
597386.2387024965421161.31664681     597465.9448     5420773.451
     597441.9324    5420403.8134     597377.4104    5420331.5317
     597393.1335    5420131.3395     597574.4756    5419951.1848
     597854.7517    5419912.8074     598081.7714    5419759.8408
     598427.0818    5419906.0503     598693.5912    5419797.6487
     598706.3272    5419673.9989     598805.7913    5419654.6798
     598981.5729    5419746.6738     599326.3572    5419741.4218
     599897.9826    5419888.6298     600287.8965     5420012.289
     600603.2217    5420175.1729     601691.3917    5421438.2026
     601948.5621    5421678.6347     602709.6031    5422228.3508
     602997.5023    5422545.3811     604028.7933    5423466.9234
     604251.6472    5423740.7625     604777.6142    5424141.3618
     605280.2617      5424704.61     605694.7374    5425052.9373
     605890.3127    5425470.3459     606173.3597    5425833.8717
     606824.0366    5426407.5418607343.2426745345426949.64970111

Type RM Length L Ch R = 1 ,43.6571 ,165.58,143.54,122.91
BEGIN DESCRIPTION:
Grand Falls Headpond
END DESCRIPTION:
XS GIS Cut Line= 2
  597695.1645036 5421183.9668831  597102.5594036 5420963.6381831
#Sta/Elev= 30
   604.2   63.59  630.73    64.2  647.73   65.73  699.71   65.64   707.7   65.17
   713.7   61.76  723.59   61.48  731.69   60.66  747.69   60.73  801.78  56.305
  805.27  56.365  808.51  57.665  821.15  56.845  831.76  57.525  844.29  57.335
  851.57  56.525  877.09  57.645  897.57  56.875  954.36  56.665  979.15  57.475
 1089.35  57.225 1113.88  58.205 1114.24   60.81 1118.53   62.67 1157.52   70.74
  1190.5   74.77  1204.5   77.22 1214.49   79.69 1229.49   81.58 1236.48   81.72
#Mann= 3 , 0 , 0
   604.2     .06       0  723.59    .035       0 1114.24     .12       0
#XS Ineff= 2 , 0
          665.19   65.92
Permanent Ineff=
       F       F
Bank Sta=723.59,1114.24
XS Rating Curve= 0 ,0
Exp/Cntr=0.3,0.1

Type RM Length L Ch R = 1 ,43.5135 ,151.21,125.11,95.9
BEGIN DESCRIPTION:
Grand Falls Headpond
END DESCRIPTION:
XS GIS Cut Line= 2
  597763.9970036 5421020.9887831  597096.9170036 5420850.6657831
#Sta/Elev= 30
     448   63.72  472.98   63.61  478.98   64.99  612.65   66.32  616.65   64.29
  621.99   63.31  627.64   60.78   670.1  57.706  696.87  56.136  699.04  56.176
   701.1  57.536  709.31  56.496  717.54  57.356  728.71  57.126   735.2  56.036
   756.3  57.086  826.14  56.046  856.92  57.196  920.59  56.446  957.21  58.436
  960.94   60.78  965.45   62.27  983.44   64.97  999.43   65.97 1021.42   66.32
 1035.41   67.87 1090.38   68.01 1109.37   70.73 1126.36   74.84 1136.36   75.61
#Mann= 3 , 0 , 0
     448     .06       0  621.99    .035       0  960.94     .12       0
#XS Ineff= 2 , 0
          612.66   66.32
Permanent Ineff=
       F       F
Bank Sta=621.99,960.94
XS Rating Curve= 0 ,0
Exp/Cntr=0.3,0.1

Type RM Length L Ch R = 1 ,43.3884 ,117.19,78.92,45.96
BEGIN DESCRIPTION:
Grand Falls Headpond
END DESCRIPTION:
XS GIS Cut Line= 3
598196.6806035985421119.79348309597703.5067035985420835.25138309
597004.9433035985420779.50268309
#Sta/Elev= 30
       0   86.11  133.85   79.25  142.84   77.42  214.76   77.92  406.55   74.93
  440.51   73.52  488.46   66.53  509.44   65.14  574.37   65.07  588.36   66.78
  599.36   65.49  636.35    65.7  645.35   62.82  656.23   62.42  710.29  56.706
   740.5  56.006  741.57  57.436  744.31  57.396  746.04  56.186  752.28  57.196
  768.28  55.596  788.91  57.066  850.34  55.516  876.36  56.986  930.56  56.026
  968.48  58.826  978.31   61.56 1041.23    67.1 1157.19   67.05 1270.15   69.97
#Mann= 3 , 0 , 0
       0    .035       0  656.23    .035       0  978.31     .12       0
Bank Sta=656.23,978.31
XS Rating Curve= 0 ,0
Exp/Cntr=0.3,0.1

Type RM Length L Ch R = 1 ,43.3095 ,77.56,50.84,23.88
BEGIN DESCRIPTION:
Grand Falls Headpond
END DESCRIPTION:
XS GIS Cut Line= 4
  597978.1346036 5420818.1539831  597617.2500036 5420716.1466831
  597306.4205036 5420759.0828831  597025.8009036 5420733.1719831
#Sta/Elev= 30
       0   81.22    7.98   80.81   23.94   78.42   40.89   74.15   63.83   71.07
  121.68   69.66  184.52   65.97   229.4    66.1  238.38   65.02   308.2   64.59
   344.1   63.28  354.08   63.67  370.04   62.19  373.03    60.7  392.01   61.16
  399.95    60.6   402.1  59.636  402.11  54.606  678.33  54.606  680.81   61.61
  717.78   63.12  754.76   65.93  758.76   65.25  765.75   65.84  799.73   65.75
  825.71   66.66  901.66   67.02  918.65   67.49  944.63   69.46  970.62   69.85
#Mann= 3 , 0 , 0
       0    .035       0  373.03    .035       0  680.81     .12       0
Bank Sta=373.03,680.81
XS Rating Curve= 0 ,0
Exp/Cntr=0.3,0.1

Type RM Length L Ch R = 6 ,43.309  ,,,
BEGIN DESCRIPTION:
Forebay Gate Structure
END DESCRIPTION:
Lateral Weir Pos= 1
Lateral Weir End=                ,                ,        ,Power Canal
Lateral Weir Distance=0
Lateral Weir TW Multiple XS=0
Lateral Weir WD=4
Lateral Weir Coef=1.45
LW OverFlow Method 2D=0
LW OverFlow Use Velocity Into 2D=0
Lateral Weir WSCriteria=-1
Lateral Weir Flap Gates= 0
Lateral Weir Hagers EQN= 0 ,,,,,
Lateral Weir SS=0.05,0.05,
Lateral Weir Type= 0
Lateral Weir Connection Pos and Dist= 3 ,
Lateral Weir SE= 2
       0  62.826      90  62.826
Lateral Weir Centerline= 0
Lateral Weir HW RS User Defined=-1
Lateral Weir HW RS Station=43.3095,0
Lateral Weir HW RS Station=43.2587,90.01
LW Gate Name Wd,H,Inv,GCoef,Exp_T,Exp_O,Exp_H,Type,WCoef,Is_Ogee,SpillHt,DesHd,#Openings
Gate #1     ,2.44,3.66,54.606,0.6,0,1,0.5, 0 ,1.67, 0 ,,, 17 ,0,0.8, 0 ,0.6,,0,0,0, 0
   16.22   19.88   23.53   27.19   30.85   34.51   38.16   41.82   45.48   50.66
   54.32   57.97   61.63   65.29   68.95    72.6   76.26
LW Gate Opening=1,Opening #1,0
LW Gate Opening=2,Opening #2,0
LW Gate Opening=3,Opening #3,0
LW Gate Opening=4,Opening #4,0
LW Gate Opening=5,Opening #5,0
LW Gate Opening=6,Opening #6,0
LW Gate Opening=7,Opening #7,0
LW Gate Opening=8,Opening #8,0
LW Gate Opening=9,Opening #9,0
LW Gate Opening=10,Opening #10,0
LW Gate Opening=11,Opening #11,0
LW Gate Opening=12,Opening #12,0
LW Gate Opening=13,Opening #13,0
LW Gate Opening=14,Opening #14,0
LW Gate Opening=15,Opening #15,0
LW Gate Opening=16,Opening #16,0
LW Gate Opening=17,Opening #17,0
LW Div RC= 0 ,False,,

Type RM Length L Ch R = 1 ,43.2587 ,255.78,14.78,12.14
BEGIN DESCRIPTION:
US of Grand Falls Main Dam
END DESCRIPTION:
XS GIS Cut Line= 3
597569.7686035985420650.02038309597308.0210035985420738.51608309
597030.5393035985420715.01628309
#Sta/Elev= 30
       0  60.906      .1  54.606   262.2  54.606  263.37  58.806  263.55  59.036
  267.33   60.87  268.32   61.84  270.32   62.44  271.32   63.96  272.31   64.57
  273.31   64.65  288.28   64.82  298.26   64.37  303.25    63.3  311.24   63.25
   331.2   64.51  348.17   65.11  362.14   64.84  372.12   65.21   382.1   65.04
  406.06    66.1  422.03   67.18  453.97   67.59  465.95   67.19   491.9   67.31
  496.89   67.53  500.88    68.1  515.85   68.55  532.82    69.6  554.78   69.66
#Mann= 3 , 0 , 0
       0    .035       0       0      .1       0  267.33     .12       0
Bank Sta=0,267.33
XS Rating Curve= 0 ,0
Exp/Cntr=0.3,0.1

Type RM Length L Ch R = 5 ,43.2577 ,,,
Node Photo=.\Photos\Grand Falls Dam.JPG
BEGIN DESCRIPTION:
Grand Falls Main Dam
END DESCRIPTION:
Node Name=GF Dam & Spillwa
IW Pilot Flow=0
#Inline Weir SE= 8
       0  60.706   244.9  60.706   244.9  63.956  246.05  63.956  246.05  60.706
   254.9  60.706   254.9  64.706   274.9  64.706
IW Dist,WD,Coef,Skew,MaxSub,Min_El,Is_Ogee,SpillHt,DesHd
0.1,4,2.1,0,0.98,, 0 ,,,3,3,
IW Gate Name Wd,H,Inv,GCoef,Exp_T,Exp_O,Exp_H,Type,WCoef,Is_Ogee,SpillHt,DesHd,#Openings
Outside Gate,6.096,3.9624,54.602,0.59,0,1,0.5, 0 ,1.67, 0 ,,, 1 ,0,0.8, 1 ,0.59,Sluice Gate Main Dam,0,0,0, 0
      11
IW Gate Opening=1,GFOG,0
IW Gate Name Wd,H,Inv,GCoef,Exp_T,Exp_O,Exp_H,Type,WCoef,Is_Ogee,SpillHt,DesHd,#Openings
Obermeyer   ,8.85,1.5,59.206,,0,1,0.5, 3 ,2.1, 0 ,,, 1 ,0,0.8, 0 ,,,0,0,0, 0
 250.475
IW Gate Opening=1,GFOB,0
IW Gate User Curve Set=Sluice Gate Main Dam
IW Gate User Curve Set Headwater=1
 61.0208
IW Gate User Curve Set Gate Opening=13
       1       2       3       4       5       6       7       8       9      10
      11      12      13
IW Gate User Curve Set Flows
 12.431124.52239 36.3022 47.742258.8424169.5744979.9667789.9909499.64698108.9349
117.7981126.2931147.2476
Inline Weir Flap Gates= 0
IW Outlet Rating Curve= 0 ,True,0,1
IW OutletRC Name=GF Power

Type RM Length L Ch R = 1 ,43.2439 ,0,11.92,18.02
BEGIN DESCRIPTION:
DS of Grand Falls Main Dam
END DESCRIPTION:
XS GIS Cut Line= 4
597556.9618035985420638.48298309597407.3939035985420690.40898309
597298.9594035995420731.87748309597032.1585035995420711.26798309
#Sta/Elev= 30
       0   57.47    .676  55.321     4.4  56.658   7.776  52.852   8.393   55.15
  14.224  54.779  14.762  56.622   17.06  53.899  54.897  55.379  77.271  52.782
  82.671  54.803  84.604  53.052  92.507  54.376   94.01  52.812  95.487  54.619
   95.84  52.905  98.308  52.495 168.656  55.313 198.699  54.731 199.537  53.187
  200.93  55.398 245.194   57.07 247.125  59.852  255.57   58.54  259.53   61.78
  260.53   63.53  268.46   64.67  303.37   63.01   420.2   67.66  542.02   69.58
#Mann= 3 , 0 , 0
       0    .035       0       0      .1       0  259.53     .12       0
Bank Sta=0,259.53
XS Rating Curve= 0 ,0
Exp/Cntr=0.3,0.1

Type RM Length L Ch R = 1 ,43.2320 ,0,81.92,129.03
XS GIS Cut Line= 3
597576.9952035985420619.82858309597273.7651035985420724.04668309
597029.2998035985420705.11098309
#Sta/Elev= 30
       0   56.95    8.17  51.706   21.82  49.706   24.83  55.546   34.03  51.906
    36.6  52.966   39.25  49.706   40.14  52.076   51.94    55.1   54.94   53.03
   65.93   54.85   77.91   53.91    87.9   54.88   93.89   52.86  107.88   52.74
  111.87   54.05  130.85   53.02  134.85   54.03   180.8   54.62  196.78    56.4
  210.76   54.53  215.76    55.3  229.74   54.16   269.7   58.81  285.68   58.49
  289.67   59.87  330.61   63.74   392.4   64.88  438.25   67.81  565.84   69.28
#Mann= 3 , 0 , 0
       0    .035       0       0      .1       0  289.67     .12       0
Bank Sta=0,289.67
XS Rating Curve= 0 ,0
Exp/Cntr=0.3,0.1

Type RM Length L Ch R = 6 ,43.231  ,,,
BEGIN DESCRIPTION:
Power Canal RCC Dam and west embankment section
END DESCRIPTION:
Lateral Weir Pos= 0
Lateral Weir End=                ,                ,        ,Power Canal
Lateral Weir Distance=0
Lateral Weir TW Multiple XS=0
Lateral Weir WD=4
Lateral Weir Coef=1.65
LW OverFlow Method 2D=0
LW OverFlow Use Velocity Into 2D=0
Lateral Weir WSCriteria=-1
Lateral Weir Flap Gates= 0
Lateral Weir Hagers EQN= 0 ,,,,,
Lateral Weir SS=0.05,0.05,
Lateral Weir Type= 0
Lateral Weir Connection Pos and Dist= 3 ,
Lateral Weir SE= 6
       0  59.806     168  59.806     168  60.716     198  63.906  431.39  63.906
     512  63.906
Lateral Weir Centerline= 0
Lateral Weir HW RS User Defined=-1
Lateral Weir HW RS Station=43.232,0
Lateral Weir HW RS Station=43.15,56
Lateral Weir HW RS Station=43.097*,112.3188
Lateral Weir HW RS Station=43.045*,167.575
Lateral Weir HW RS Station=42.9919,224
Lateral Weir HW RS Station=42.926*,278.5
Lateral Weir HW RS Station=42.8601,333
Lateral Weir HW RS Station=42.8015,342
Lateral Weir HW RS Station=42.749*,384.554
Lateral Weir HW RS Station=42.697*,426.7026
Lateral Weir HW RS Station=42.645*,468.8513
Lateral Weir HW RS Station=42.593,511
Lateral Weir HW RS Station=42.538*,530
LW Gate Name Wd,H,Inv,GCoef,Exp_T,Exp_O,Exp_H,Type,WCoef,Is_Ogee,SpillHt,DesHd,#Openings
Inside Gate ,4.572,2.1336,54.602,0.59,0,1,0.5, 0 ,1.67, 0 ,,, 1 ,0,0.8, 1 ,0.59,,0,0,0, 0
      10
LW Gate Opening=1,GFIG,0
LW Gate Name Wd,H,Inv,GCoef,Exp_T,Exp_O,Exp_H,Type,WCoef,Is_Ogee,SpillHt,DesHd,#Openings
RCC Fboards ,168,0.9,59.806,,0,1,0.5, 3 ,1.8, 0 ,,, 1 ,0,0.8, 0 ,,,0,0,0, 0
      84
LW Gate Opening=1,GFRCCFB,0
LW Div RC= 0 ,False,,

Type RM Length L Ch R = 1 ,43.1500 ,56.333,105.41,111.457
XS GIS Cut Line= 2
597571.8794035995420564.08708309597025.4067035985420630.16758309
#Sta/Elev= 30
       0   54.97    5.99   52.16   10.99   52.75   13.99    50.6   24.98   50.82
   30.97   53.07   40.96   52.24   42.96    50.5   51.95   51.39   56.94   53.78
   67.93   52.54   85.91    54.8   102.9   51.27  113.89   52.68  116.88    49.8
  151.85   51.97  165.84   49.86  175.83   51.48  177.82   49.52  190.81   46.93
   205.8   47.64  210.79   49.36  213.79   51.33  216.78   56.29  223.78   59.85
  257.74   61.02  269.73   63.82  363.64   65.55  414.59   64.48  550.45   68.05
#Mann= 3 , 0 , 0
       0    .035       0       0      .1       0  216.78     .12       0
Bank Sta=0,216.78
XS Rating Curve= 0 ,0
Exp/Cntr=0.3,0.1

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
Type RM Length L Ch R = 1 ,42.9919 ,159.645,115.34,119.86
XS GIS Cut Line= 2
597531.1858035985420409.68748309596992.9203035985420476.67608309
#Sta/Elev= 30
       0   52.98    8.39   49.98   13.98   48.94   17.98   46.98   25.97   44.95
   54.94   44.75   56.94   43.82   79.91   42.49   85.91   42.64  104.89   46.58
  118.87   43.75  124.87    45.6  160.71   45.58  167.82   45.69  173.81   47.17
  178.81   45.86   185.8   46.71  202.78   46.48  223.76   47.04  230.75   47.85
  233.75   48.65  256.72    64.4  260.72   66.07  288.69   66.06  307.67   64.33
   374.6   64.51  394.58   65.18  406.56   67.03  428.54   64.91  542.42    65.4
#Mann= 3 , 0 , 0
       0    .035       0    8.39      .1       0  160.71     .12       0
Bank Sta=8.39,160.71
XS Rating Curve= 0 ,0
Exp/Cntr=0.3,0.1

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
Type RM Length L Ch R = 1 ,42.8601 ,54.26,58.64,95.11
XS GIS Cut Line= 3
597495.0681035985420306.46288309597212.0706035985420331.30568309
597193.7150035985420278.68958309
#Sta/Elev= 30
       0      54   12.96   53.42   22.93    49.6   35.88   47.81   41.87   45.13
   47.85   44.17    62.8   43.72   77.75   44.67   85.72    42.1   88.71   39.39
    91.7   37.86   97.69   37.66  107.65    35.5  108.91   34.38  110.64   32.19
  114.63   31.54  131.58   31.65  139.55   32.98  141.54   34.79  145.53   44.26
  146.01   44.55  152.51   44.58  159.49   46.08  167.46   45.78  213.31   52.82
  219.29   55.07  233.25   62.74  238.23   64.05  275.11   65.61  339.81   70.57
#Mann= 3 , 0 , 0
       0      .1       0  108.91      .1       0  146.01     .12       0
Bank Sta=108.91,146.01
XS Rating Curve= 0 ,0
Exp/Cntr=0.3,0.1

Type RM Length L Ch R = 1 ,42.8015 ,102.183,117.272,109.268
XS GIS Cut Line= 2
597492.4103035985420297.95878309597074.4635035985420142.98428309
#Sta/Elev= 30
       0   54.23   16.99   52.49   27.98   49.79   45.97   48.61   49.97    46.8
   52.97   44.05   61.97   41.77   78.96   41.98   81.95   43.65   85.95   43.68
   92.95   45.64   97.23    44.8   98.95    41.7   99.94   37.92  100.94   35.87
  103.94   35.16  107.94   31.59 115.385  31.206  166.91    31.6  173.67   33.92
   177.9   34.37   182.9   36.88  196.89   52.19  200.89    55.1  227.87   60.45
  240.87   62.28  312.83    69.6   355.8   69.08  402.78   70.45  445.75   70.46
#Mann= 3 , 0 , 0
       0      .1       0   97.23      .1       0  173.67     .12       0
Bank Sta=97.23,173.67
XS Rating Curve= 0 ,0
Exp/Cntr=0.3,0.1

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
Type RM Length L Ch R = 1 ,42.5930 ,94.2,110.187,126.55
XS GIS Cut Line= 3
597540.0600035985420134.24288309597136.0700035985419954.32478309
597055.4412035985420050.61358309
#Sta/Elev= 30
       0   48.71    8.98   51.55   28.95   49.09   38.93   55.51   62.89   54.98
   76.87   51.22   78.86   47.84   81.86      39   86.99    33.2   88.85   29.47
   90.84   28.02  101.64  26.207   114.8   29.81   117.8   28.61  129.78    32.7
  134.13   31.28  141.76   34.41  166.71   35.77   173.7   39.06  178.69   38.85
  198.66   51.93  203.65   50.37  216.63   54.69   232.6   54.02  244.58    49.4
  262.55   56.11  279.52   57.42   485.1   62.77  540.92   69.46  567.83   70.25
#Mann= 3 , 0 , 0
       0     .08       0   86.99      .1       0  134.13     .12       0
Bank Sta=86.99,134.13
XS Rating Curve= 0 ,0
Exp/Cntr=0.3,0.1

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
Type RM Length L Ch R = 1 ,42.4277 ,122.945,136.96,163.235
BEGIN DESCRIPTION:
Grand Falls Powerhouse
END DESCRIPTION:
XS GIS Cut Line= 2
597612.5543035995420143.22608309597357.4101035995419438.13158309
#Sta/Elev= 30
       0   52.14   58.99   51.62   74.98   49.41   82.98    43.6   88.98    42.8
   91.98   44.95   97.98   45.03  104.98   41.51  118.97   41.17  133.97   33.08
  134.97   31.31  135.56  25.707 139.829  25.707     140   25.65     200   25.65
  225.14   28.57  243.95   34.39  248.95   30.49  255.94   30.24  267.94   37.57
  281.94   32.74  299.93   32.23  307.93   33.71  322.93   40.16  369.92   47.11
  426.91   47.09  519.89   58.97  566.88   58.23  678.85   64.18  749.84   64.54
#Mann= 3 , 0 , 0
       0     .08       0 139.829    .035       0  225.14     .12       0
Bank Sta=139.829,225.14
XS Rating Curve= 0 ,0
Exp/Cntr=0.3,0.1

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
Type RM Length L Ch R = 1 ,42.2908 ,102.61,105.315,118.92
XS GIS Cut Line= 2
597687.2405035985420126.97068309597644.8885035985419425.34598309
#Sta/Elev= 30
       0   52.83   67.99   51.64   73.99   50.42   78.99   46.74   86.99   44.32
  104.99   44.05  116.98   36.48  127.98   32.94  153.98   31.46  160.55   28.45
     171    24.7     251    24.7  254.75  26.087  272.67   27.16  281.96   31.18
  284.96   38.08  287.96   40.66  307.96   38.09  319.95   40.72  375.95   46.37
  435.94   47.23  456.94   48.61  513.93   57.31  519.93   60.69  558.92   60.62
  564.92   62.74  577.92   63.87  585.92   66.34  619.91   69.55   702.9   73.13
#Mann= 3 , 0 , 0
       0     .08       0  160.55      .1       0  272.67     .12       0
Bank Sta=160.55,272.67
XS Rating Curve= 0 ,0
Exp/Cntr=0.3,0.1

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
Type RM Length L Ch R = 1 ,42.1704 ,99.05,82.24,54.4
XS GIS Cut Line= 3
597775.8355035995420082.58128309597808.5226035985419810.51958309
597692.5833035995419573.53828309
#Sta/Elev= 30
       0   53.99   59.79   53.31   66.76   51.35   75.73   51.61   91.67   43.53
  100.64   44.02   112.6      42  123.57   31.01  131.53   25.32     137    23.3
     187    23.3  190.75  25.042  198.29   25.47  215.93   32.24  232.17   36.51
  246.12   42.39  259.07   43.26  270.03   48.09  283.01    44.3  290.01   46.65
     303   44.63  326.98   49.87  425.92   50.31   448.9   52.79  459.89   57.57
  470.89   58.97  489.87   60.47  503.86   57.93  522.85   59.15  537.84   63.56
#Mann= 3 , 0 , 0
       0     .08       0  123.57      .1       0  215.93     .12       0
Bank Sta=123.57,215.93
XS Rating Curve= 0 ,0
Exp/Cntr=0.3,0.1

Type RM Length L Ch R = 1 ,42.0882 ,39.86,40.01,40.58
BEGIN DESCRIPTION:
US Mill Bridge
END DESCRIPTION:
XS GIS Cut Line= 2
597955.2319035995420067.01388309597690.6361035985419542.94588309
#Sta/Elev= 30
       0   54.97  122.81   51.67  133.79   50.28  142.78   44.56  147.77   43.38
  151.76   33.03  153.76   32.92  156.75   26.58  158.75   25.28 192.265  22.712
  224.65    24.9  227.74   26.31  232.63   29.97  237.63   38.68  244.62   42.76
  265.58   42.48  279.56   44.97  287.55   44.11  294.54   46.56  308.51   44.28
  340.46   49.29  430.32   49.84  455.28   51.28  497.22   58.37   505.2   56.59
  528.17    57.9  538.15   62.62  568.11   66.84   574.1   70.43  587.08   72.19
#Mann= 3 , 0 , 0
       0     .08       0  158.75    .035       0  227.74     .12       0
Bank Sta=158.75,227.74
XS Rating Curve= 0 ,0
Exp/Cntr=0.3,0.1

Type RM Length L Ch R = 1 ,42.0481 ,69.91,67.89,65.71
BEGIN DESCRIPTION:
DS Mill Bridge
END DESCRIPTION:
XS GIS Cut Line= 2
597997.0352035985420060.35468309597728.8329035985419533.00958309
#Sta/Elev= 30
       0   55.05   64.96   51.33  108.93   49.98  122.92   50.54  126.92   49.63
   159.9    49.1   164.9   47.41  167.89   45.05  168.89   43.03  170.89   33.66
  171.89   31.27  179.89   24.89 206.025  22.712  227.86   25.71  229.86   28.05
  231.98   33.35  232.85   34.94  235.85   43.77  238.85   46.43  239.85   48.12
  241.85    49.1  304.81   48.22  420.74   50.27   477.7   52.76  486.69   53.77
  495.69   56.41  517.67    58.8  560.65   66.29  580.64   68.66  591.63   68.69
#Mann= 3 , 0 , 0
       0     .12       0  170.89    .035       0  231.98     .12       0
Bank Sta=170.89,231.98
XS Rating Curve= 0 ,0
Exp/Cntr=0.3,0.1

Type RM Length L Ch R = 1 ,41.9803 ,105.17,113.56,170.98
XS GIS Cut Line= 2
598131.3099035985420112.89648309597740.0376035985419490.01148309
#Sta/Elev= 30
       0   54.93   62.96   53.47   76.96   51.27  242.86   53.11  265.85   51.41
  288.84   47.66  291.83   43.82   297.3   33.82  303.83    25.6 332.335  22.712
  354.62   24.94   358.8   25.92  364.79   30.31  373.79   39.25  400.77   40.45
  408.77   43.11  427.76   46.02  459.74   47.92  485.72   46.06  493.72   48.96
  501.71   49.84   535.7   49.28  549.69    47.3  585.67   51.31  601.66   55.69
  618.65   54.94  637.64   56.32  684.61   67.61   704.6   65.26  735.58   66.78
#Mann= 3 , 0 , 0
       0     .12       0   297.3    .035       0  354.62     .12       0
Bank Sta=297.3,354.62
XS Rating Curve= 0 ,0
Exp/Cntr=0.3,0.1

Type RM Length L Ch R = 1 ,41.8667 ,94.84,121.425,152.8
XS GIS Cut Line= 2
598145.1294035995420109.78868309597982.5971035995419513.98098309
#Sta/Elev= 30
       0   54.75   75.95   51.35   79.95   52.78   86.94   52.93   92.94   50.84
   144.9   49.08   149.9    47.7  158.89   50.55  166.89   51.27  185.87   48.53
  209.86   48.19  229.84   45.06  253.83   44.77  265.82   42.55  270.82   36.97
  279.81   29.36  284.81   26.14  287.96   25.52  294.93   23.35  365.47    23.3
  421.85   23.34  439.22   28.07   446.7   29.23  462.68   38.24  505.66   40.81
  565.61    51.4  573.61   54.73  594.59   56.38  602.59   60.15  617.58   55.88
#Mann= 3 , 0 , 0
       0     .12       0  287.96    .035       0  439.22     .12       0
Bank Sta=287.96,439.22
XS Rating Curve= 0 ,0
Exp/Cntr=0.3,0.1

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
Type RM Length L Ch R = 1 ,41.6238 ,150.015,113.19,92.86
XS GIS Cut Line= 2
  598156.4052036 5420113.0567831  598336.5925036 5419668.8636831
#Sta/Elev= 30
       0   55.04   12.98   54.24   18.97   53.23   35.95   53.14   63.91   51.85
  105.86   45.16  133.82   44.33  157.79   42.39  175.76   42.51  181.75   38.66
  185.75   38.83  198.73   36.74  208.72   36.37   218.7   30.38  225.31   27.15
  234.68   23.93 298.275  20.914  361.51   24.76  364.51   27.67   365.5   29.54
   366.5   32.55   367.5   34.34   371.5    39.5  375.49   40.25  380.76   39.84
  388.47   40.14  407.45   45.86   443.4   50.58  455.38   54.14  479.35    53.6
#Mann= 3 , 0 , 0
       0     .12       0  225.31    .035       0  380.76     .12       0
Bank Sta=225.31,380.76
XS Rating Curve= 0 ,0
Exp/Cntr=0.3,0.1

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
Type RM Length L Ch R = 1 ,41.3975 ,123.69,82.54,74.28
XS GIS Cut Line= 3
  598528.7382036 5420435.1340831  598524.4723036 5420116.4904831
  598434.5741036 5419681.6617831
#Sta/Elev= 30
       0   70.96   10.99   70.66   15.98    69.2   41.96      69   55.94   66.72
   81.92   59.03  103.89   59.17  139.86   56.45   287.7   51.89  318.67    50.5
  326.66   47.89  386.52   46.13  400.49   38.57  412.47   37.21  416.46   32.96
  424.44   27.73  438.41   23.27  446.16   22.86  480.27  20.914  523.13  22.214
  565.99  20.914  606.19   23.74  611.03   26.14  618.02   32.55  619.01   34.49
  620.01   38.32     627   40.41  679.88   46.42  708.82   48.66   762.7   50.15
#Mann= 3 , 0 , 0
       0     .12       0  446.16    .035       0  606.19     .12       0
Bank Sta=446.16,606.19
XS Rating Curve= 0 ,0
Exp/Cntr=0.3,0.1

Type RM Length L Ch R = 1 ,41.3149 ,99.285,88.355,80.53
XS GIS Cut Line= 3
  598663.5854036 5420441.1382831  598662.2569036 5420130.2724831
  598477.5198036 5419674.8176831
#Sta/Elev= 30
       0   59.71   50.98   57.01   68.97   57.34   83.96   55.79  170.93   53.77
   237.9   53.96  303.87    51.2  310.87   49.53  320.86   49.52  330.85   46.52
  342.84   46.98   376.8   45.44  384.79   41.36  511.66   37.62  520.65   34.67
  553.45   28.47  561.61   26.63  563.61   24.41  593.99   20.19  628.03   20.21
  638.53   22.45  640.53   23.76  642.53   27.98  645.52      36  650.52   38.32
   664.5   39.04   671.5   38.34  680.49   40.78  742.42   47.81  802.36   50.05
#Mann= 3 , 0 , 0
       0     .12       0  553.45    .035       0  642.53     .12       0
Bank Sta=553.45,642.53
XS Rating Curve= 0 ,0
Exp/Cntr=0.3,0.1

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
Type RM Length L Ch R = 1 ,41.1382 ,63.25,126.28,148.07
XS GIS Cut Line= 3
  598800.5850036 5420456.0698831  598795.8666036 5419849.6393831
  598489.4724036 5419610.6914831
#Sta/Elev= 30
       0   53.32   54.95   51.26  156.86      52  243.78   50.04  314.71   52.15
  363.67   44.46  383.65   45.36  387.65   43.27  412.62   42.23  508.54   41.37
  533.52    42.8   546.5   38.68  559.49   40.88  563.49    39.2  588.47   41.42
  618.44   39.53  636.41   40.95   645.4   38.17   651.4   28.57  655.39    25.7
  676.79   22.29  683.36   23.41  700.87    19.3  736.68   19.31  758.51    24.4
  777.25   34.34  837.18    28.9  890.12   39.63  919.09   47.62     995   50.06
#Mann= 3 , 0 , 0
       0     .12       0  676.79    .035       0  758.51     .12       0
Bank Sta=676.79,758.51
XS Rating Curve= 0 ,0
Exp/Cntr=0.3,0.1

Type RM Length L Ch R = 1 ,41.0119 ,22.93,94.61,179.55
XS GIS Cut Line= 4
  598905.8685036 5420527.1683831  598858.6945036 5419869.8341831
  598539.9867036 5419427.5964831  598454.2653036 5419405.6642831
#Sta/Elev= 30
       0   54.99  145.78   50.67  378.44   51.69  505.25   39.93  564.17   43.82
  570.16   40.81  621.08   41.67  640.05   31.39  731.91   32.95  742.89   27.07
  754.87   31.55  783.07   25.31  821.82  18.745  841.73   24.12  845.72   21.05
  849.71   31.45   855.7    36.7  867.68   32.48  868.68   31.22  870.68   20.58
  901.83  17.715  935.57   21.18  947.55   27.74  961.53   25.22  965.52   20.07
  979.56   20.38 1034.41   28.26 1088.32   28.85 1174.18   44.19 1292.62   45.07
#Mann= 3 , 0 , 0
       0     .12       0  783.07    .035       0  979.56     .12       0
Bank Sta=783.07,979.56
XS Rating Curve= 0 ,0
Exp/Cntr=0.3,0.1

Type RM Length L Ch R = 1 ,40.9173 ,104.51,124.65,154.26
XS GIS Cut Line= 4
  599026.1086036 5420540.6695831  598902.4502036 5419926.0542831
  598790.4353036 5419769.2360831  598869.5036036 5419034.6033831
#Sta/Elev= 30
       0   53.22   94.99      51  312.97   52.06  536.94   43.05  573.94   44.78
  596.94   40.45  604.93   43.75  638.91   44.79   646.9   41.87   650.9   37.43
  677.86   31.46  767.73   32.51  772.72   32.01  781.71   26.38  801.68   29.57
  841.38   20.32  892.32   18.08  992.62    19.3 1002.62   23.53 1007.62   29.14
 1010.45   35.17 1013.61   38.83 1029.61   37.08 1041.61   29.61 1054.61    28.4
  1108.6   30.49 1299.58   27.95 1362.57   30.33 1404.56   37.75 1558.54   39.36
#Mann= 3 , 0 , 0
       0     .12       0  841.38    .035       0 1010.45     .12       0
Bank Sta=841.38,1010.45
XS Rating Curve= 0 ,0
Exp/Cntr=0.3,0.1

Type RM Length L Ch R = 1 ,40.7927 ,135.24,97.35,89.19
XS GIS Cut Line= 5
  599071.2521036 5420532.4645831  598959.0884036 5419969.0653831
  598863.4854036 5419835.5306831  598920.5291036 5419682.8368831
  598977.4507036 5419085.5791831
#Sta/Elev= 30
       0   53.04   425.6   48.65  462.56   45.29   529.5   44.84  572.46   40.67
  599.34   43.33  615.26   38.08  627.21   40.61  688.92    32.6  747.63   29.03
  786.39   28.67   796.8   31.28  806.27   28.57  808.26   19.59  810.24   19.02
 853.695  17.016  913.63   21.08  923.68    23.7  950.68   22.46  973.68   27.84
 1018.68   29.73 1204.66   28.96 1219.66   30.84 1238.66   38.04 1258.66   37.25
 1275.65   29.44 1327.65   30.66 1353.65   36.37 1390.64   37.91 1501.64   36.48
#Mann= 3 , 0 , 0
       0     .12       0   796.8    .045       0  913.63     .12       0
Bank Sta=796.8,913.63
XS Rating Curve= 0 ,0
Exp/Cntr=0.3,0.1

Type RM Length L Ch R = 1 ,40.6953 ,368.69,407.83,456.42
BEGIN DESCRIPTION:
R13 (RIS 2013)
END DESCRIPTION:
XS GIS Cut Line= 3
  599099.2065036 5420529.6327831  598954.0399036 5419398.3266831
  598982.9888036 5419112.7675831
#Sta/Elev= 30
       0   53.31  110.96   52.03  139.95   48.65  316.88   47.67  387.86   48.44
  418.85   52.89  426.84   48.22   555.8   46.43  575.79   41.36  593.78   42.91
  606.78   38.29  642.76    37.6  677.75   32.37  695.75   23.21   706.6   20.92
  804.92  12.946  818.38  13.676  833.05  18.496  928.07   18.84  947.65   21.49
  965.65   28.92 1151.55   28.99 1167.49   30.41 1178.46   36.48 1191.41   37.54
 1213.34   37.13 1226.29   29.71 1277.12   30.61 1335.92   37.86 1427.61   35.65
#Mann= 3 , 0 , 0
       0     .12       0   706.6    .045       0  928.07     .12       0
Bank Sta=706.6,928.07
XS Rating Curve= 0 ,0
Exp/Cntr=0.3,0.1

Type RM Length L Ch R = 1 ,40.2875 ,574.92,574.64,644.45
BEGIN DESCRIPTION:
R14 (RIS 2013)
END DESCRIPTION:
XS GIS Cut Line= 4
599214.1084035985420543.04368309599438.2531035985419613.21718309
599419.7029035995419515.35288309599491.4356035985419090.56948309
#Sta/Elev= 30
       0   51.91  215.88   47.79  293.83   57.33  380.79   59.02  413.77   56.27
  436.75   48.59  477.73   40.75  499.72   41.15  510.71   37.74   525.7   38.98
   533.7   36.67  565.68   35.16  598.66    19.8  669.01   19.55  712.83  15.647
  865.61  15.777  922.84    19.7  959.46    23.7 1031.17   24.78 1046.11   35.38
  1050.1   36.22 1090.06   35.97 1125.04   39.57 1148.03   34.88 1166.02   38.93
 1326.94   35.88 1369.92   39.42  1394.9   45.02 1441.88   45.31 1486.86   50.13
#Mann= 3 , 0 , 0
       0     .12       0  669.01    .045       0  922.84     .12       0
Bank Sta=669.01,922.84
XS Rating Curve= 0 ,0
Exp/Cntr=0.3,0.1

Type RM Length L Ch R = 1 ,39.7129 ,581.88,619.1,724.22
BEGIN DESCRIPTION:
Gorge Park - R15 (RIS 2013)
END DESCRIPTION:
XS GIS Cut Line= 2
599798.9278035985420261.30898309600162.7547035985419452.58748309
#Sta/Elev= 30
       0   37.66       6    35.1   22.99   32.75   89.98   30.01  120.97   29.69
  123.97    29.3  128.97   26.67  141.97   22.93   190.5   21.37  196.95   18.91
  219.12  18.048  238.91  16.138  271.27  15.928  402.76  16.838  459.76  18.108
   541.6  16.798  591.18  18.138  618.51   20.77  628.85   22.78  640.85   20.44
  689.84   22.57  733.83   21.87  743.83   26.48  752.82   32.23  760.82   31.73
  795.81   38.51   837.8   40.63   867.8   47.29   879.8      48  886.79   51.41
#Mann= 3 , 0 , 0
       0     .12       0   190.5    .045       0  618.51     .12       0
Bank Sta=190.5,618.51
XS Rating Curve= 0 ,0
Exp/Cntr=0.3,0.1
