HEC-RAS study Unsteady_RAS.prj: Unsteady_RAS

--- Unsteady_RAS.g01 (geometry) --- (continued)

Type RM Length L Ch R = 1 ,126.7103,47.22,47.56,47.15
BEGIN DESCRIPTION:
DS of Exploits Bridge
END DESCRIPTION:
XS GIS Cut Line= 6
     530712.6945    5401840.7123     530750.1104    5401634.2396
     530742.7448    5401318.4032     530755.5081    5400671.5793
     530622.7564    5400341.2659     530510.0752    5399877.1315
#Sta/Elev= 30
       0  197.49   28.98   197.9   70.94  192.88   88.93  193.14  109.91  187.91
  290.65  180.65   489.9  165.66  528.78  164.25  631.73  166.75  709.66  158.55
  717.63  155.93  817.74   149.2 823.845 148.429  826.87 145.225 915.866 145.225
  916.98 147.225 1039.41  149.72 1237.99  157.53 1314.71  165.98 1322.67  164.61
 1375.41  167.13 1394.32  165.53 1492.06  173.55 1564.42  171.57 1626.37  173.13
 1731.28  169.26  1826.2  172.53 1893.15  170.18 1934.12  175.47 2007.06  173.72
#Mann= 3 , 0 , 0
       0     .12       0  826.87    .035       0  916.98     .12       0
Bank Sta=826.87,916.98
XS Rating Curve= 0 ,0
Exp/Cntr=0.3,0.1

Type RM Length L Ch R = 1 ,126.6627,636.49,615.55,614.09
XS GIS Cut Line= 3
     530777.8506    5401823.3022     530804.9257    5400768.2052
     530546.9935     5399862.792
#Sta/Elev= 30
       0   196.8   48.97  194.05   56.97  190.99   81.96  188.91  290.85  180.26
  492.74  164.01  552.71   162.7   567.7  165.74  589.69  166.08  654.66  157.37
  692.64  155.76   771.6  147.72  785.59  148.56  795.01 145.225  891.13 145.225
  894.53   148.1  903.53  148.66 1006.47     150 1241.33  158.52 1265.32  161.02
 1277.31  158.99 1335.28  163.03 1362.26  162.29 1446.21  170.22 1498.18  172.28
 1588.12  170.03  1635.1  164.78 1672.07  164.43 1810.99  173.03 1996.88  175.14
#Mann= 3 , 0 , 0
       0     .12       0  795.01    .035       0  891.13     .12       0
Bank Sta=795.01,891.13
XS Rating Curve= 0 ,0
Exp/Cntr=0.3,0.1

Type RM Length L Ch R = 1 ,126.0472,263.67,275.39,451.09
XS GIS Cut Line= 6
     531431.9082     5401732.948     531423.0495    5401069.4261
     531421.9701    5400988.5859     531405.4493    5400889.6454
     531363.2926    5400637.1753     531167.2506    5399463.1203
#Sta/Elev= 30
       0  183.85  131.92  174.21  205.87  173.36  352.78  164.34  619.61   155.4
  673.56   150.9  709.49  152.93  752.37  146.66 753.848 144.625  908.26 144.625
  912.73  146.92  998.72  149.67 1090.71  150.55 1197.65  149.32 1223.63  151.37
  1278.6   152.3 1354.55   150.3 1879.23  188.18 2091.11  199.07 2093.11  202.29
  2098.1  203.72 2134.08  205.39 2136.08  207.18 2154.07  206.82 2156.07  208.75
 2193.05  208.75 2195.05  210.37 2213.04  210.37 2234.03  212.61    2291  213.72
#Mann= 3 , 0 , 0
       0     .12       0  752.37    .035       0  908.26     .12       0
Bank Sta=752.37,908.26
XS Rating Curve= 0 ,0
Exp/Cntr=0.3,0.1

Type RM Length L Ch R = 1 ,125.7718,856.73,915.26,1015.11
XS GIS Cut Line= 6
     531651.5385    5401693.5439     531671.3391    5401103.2408
     531678.8104    5400880.4983     531682.8283    5400760.7109
     531697.0695    5400656.0296     531823.3568     5399727.734
#Sta/Elev= 30
       0   179.7  180.89  170.63   324.8  167.88  468.71  158.46  559.65  155.48
  578.64  153.19 615.273 144.401 653.281 144.382   654.6  146.69  762.54  145.82
 769.305 143.874 795.287 143.894  800.51  145.73  808.51  147.41   898.4  148.01
 1047.01  147.38    1069  145.141092.522 143.7771163.047 144.022 1165.99  146.88
 1174.99  148.79 1277.97  162.18 1495.94  182.41 1531.93     183 1540.93  185.44
 1577.93  186.62 1663.91  194.71 1672.91  193.54 1722.91  199.44 1975.87  213.02
#Mann= 7 ,-1 , 0
       0     .12       0 615.273    .035       0   654.6     .12       0
  762.54    .035       0  800.51     .12       0    1069    .035       0
1163.047     .12       0
Bank Sta=615.273,1163.047
XS Rating Curve= 0 ,0
Exp/Cntr=0.3,0.1

Type RM Length L Ch R = 1 ,124.8565,379.59,352.29,333.1
XS GIS Cut Line= 6
     532300.8986    5401888.1507     532527.3127    5401162.0206
     532551.2177    5401105.3231     532619.6728    5400942.9625
     532868.0471    5400353.8708     533049.1264    5399778.5236
#Sta/Elev= 30
       0  180.84   57.98  178.25  137.94  171.34   224.9  171.99  325.86  168.26
  609.74  153.03  676.69   144.8  727.64  146.78  737.06 144.727  808.31 142.507
  883.01 144.727  883.87  146.32  886.85  146.93   943.6  149.39 1019.33   149.9
  1045.3  151.42 1064.28  154.15 1107.23  155.48 1127.21   159.3 1164.17  158.78
 1225.11  165.83 1282.05   168.9 1346.98  176.73 1602.71   190.5 1660.64  192.17
 1724.56  196.15 1872.35  198.67 1971.21  202.15 2134.99   211.1 2240.85  214.35
#Mann= 3 , 0 , 0
       0     .12       0  737.06    .035       0  883.01     .12       0
Bank Sta=737.06,883.01
XS Rating Curve= 0 ,0
Exp/Cntr=0.3,0.1

Type RM Length L Ch R = 1 ,124.5042,337.4,401.89,491.22
XS GIS Cut Line= 6
     532488.5325     5402103.292     532820.9539    5401459.7091
     532859.8394    5401384.4248     532882.2562    5401127.6003
     532909.2417    5401065.9085     533412.4003    5399915.6244
#Sta/Elev= 30
       0  182.83   111.9  180.38  154.86  176.59  179.84  175.96  190.83  173.76
  587.49   154.7     835  149.16   862.9  147.52  874.85  145.14  878.09 142.728
 997.775 142.728  997.91 144.881 1002.27  145.93 1089.68  144.86 1352.16  166.41
 1427.13  170.72 1452.12  169.89 1568.08  171.24 1824.99  185.62 1913.96  189.27
 1966.94  190.06 2025.92  193.46  2063.9  193.33 2082.89  194.97 2185.85  194.42
 2261.82  196.53  2318.8  195.86 2343.79  193.85 2356.78  194.98 2389.77  193.51
#Mann= 3 , 0 , 0
       0     .12       0  878.09    .035       0  997.91     .12       0
Bank Sta=878.09,997.91
XS Rating Curve= 0 ,0
Exp/Cntr=0.3,0.1

Type RM Length L Ch R = 1 ,124.1023,533.43,530.75,532.18
BEGIN DESCRIPTION:
E37 (SEM 2016)
END DESCRIPTION:
XS GIS Cut Line= 6
     532505.7291    5402099.0737     532987.0839    5401619.7142
     533081.4557    5401525.7334     533222.4342    5401426.0061
     533539.2532    5400988.9358     533553.4569    5399906.6829
#Sta/Elev= 30
       0  182.28  115.89   180.8  160.84  174.66   303.7  164.66   400.6  161.71
  519.49  154.68  683.31  150.45  716.11   150.8  772.76  154.79  802.57  150.56
   818.5 145.409 820.455 142.252  857.68 140.115 925.866 143.056  937.91  145.47
 1100.74  148.54 1170.62  151.64 1221.54  155.94 1282.43   155.7 1355.31  159.47
  1417.2  159.23 1612.96  165.51 1864.81  167.82 1899.79  171.54 1940.77  169.71
 1991.74  171.13 2254.56  182.85 2421.44  183.38 2505.38  185.25 2607.31  184.69
#Mann= 3 , 0 , 0
       0     .12       0   818.5    .035       0  937.91     .12       0
Bank Sta=818.5,937.91
XS Rating Curve= 0 ,0
Exp/Cntr=0.3,0.1

Type RM Length L Ch R = 1 ,123.5716,239.58,203.22,170.46
BEGIN DESCRIPTION:
Harpoon Brook
END DESCRIPTION:
XS GIS Cut Line= 6
     532796.3526    5402351.7543     533234.9884    5402054.2969
     533558.6234    5401834.8259     533723.0683    5401640.1773
     534261.7597     5401228.239      534271.281     5401228.364
#Sta/Elev= 30
       0  179.81      48  174.71  416.99  156.63  440.99  154.37  606.64  149.49
  620.58  148.23   638.5  144.57 685.855 143.337  764.16  143.88  771.15  148.65
  779.15  149.01  990.52   150.5 1043.32  153.27 1097.12  154.04 1247.74  152.71
 1298.68  157.89 1324.64  156.05 1354.61  155.96 1506.41  160.59 1551.36   163.2
 1657.22  163.13 1734.12  171.11 1761.09  172.22 1797.04  171.99 1817.02  170.21
 1824.01  171.65 1837.99  171.69 1845.98  169.52 1850.97   171.1 1863.49  171.14
#Mann= 3 , 0 , 0
       0     .12       0   638.5    .035       0  764.16     .12       0
Bank Sta=638.5,764.16
XS Rating Curve= 0 ,0
Exp/Cntr=0.3,0.1

Type RM Length L Ch R = 1 ,123.3684,254.4,206.7,170.81
XS GIS Cut Line= 6
     533088.7417    5403292.0131     533378.7206    5402822.0506
     533494.1975    5402148.2367     533664.7161    5401818.1051
     533689.6226    5401769.8849     534299.0118    5401292.2143
#Sta/Elev= 30
       0  182.35   211.7  180.53   425.4  175.65  451.37  173.53  617.14  170.99
   865.8  159.95 1096.49  154.62 1177.17  150.17  1191.1     147 1211.99  145.36
1221.809 142.151 1247.39 142.1271354.721 142.172 1355.71  143.62  1359.7  146.18
 1386.67  147.56 1445.61  145.51 1513.53  149.16 1674.69  153.65 1845.53  152.37
  1878.5  155.87 1980.41  158.93 2016.38  162.55 2060.34  161.59 2156.25  165.82
 2183.22   163.2 2216.19  163.39 2269.14  171.66 2336.07  173.75 2435.97  172.12
#Mann= 3 , 0 , 0
       0     .12       01221.809    .035       0 1355.71     .12       0
Bank Sta=1221.809,1355.71
XS Rating Curve= 0 ,0
Exp/Cntr=0.3,0.1

Type RM Length L Ch R = 1 ,123.1617,264.8,285.33,341.35
XS GIS Cut Line= 6
     533367.3243    5403349.6339     533641.1778    5402850.9695
     533735.0284    5402179.9669     533699.9013    5401954.1298
     533785.1272    5401748.9184     534333.0067    5401362.4953
#Sta/Elev= 30
       0  180.06  198.97   177.6  409.94  167.86  417.94  168.82  510.92  166.39
  694.77  159.04   835.6  157.57 1023.37  158.82 1218.67  157.41 1244.47  146.89
1303.947 142.265 1394.82 142.048 1400.36  146.57 1405.34  147.13 1458.08  143.88
 1513.79  144.55 1621.31   153.1 1696.21  153.82 1793.13  152.31 1836.09  156.02
 1892.04  156.01    1945  162.08 2048.91  163.46 2082.89  166.23 2105.87  164.42
 2137.85   164.6 2162.83  168.41 2237.77  173.54 2298.72  174.97 2367.67  173.12
#Mann= 3 , 0 , 0
       0     .12       01303.947    .035       0 1394.82     .12       0
Bank Sta=1303.947,1394.82
XS Rating Curve= 0 ,0
Exp/Cntr=0.3,0.1

Type RM Length L Ch R = 1 ,122.8763,427.62,460.15,513.31
XS GIS Cut Line= 6
     533555.9164    5403491.7797     533801.2509    5403177.0837
      533942.971    5402315.2208     534014.0772    5401882.7897
     534060.0289    5401603.3343     534329.0414    5401422.7552
#Sta/Elev= 30
       0  183.21  218.47  177.51  299.27  171.72  474.98  162.98  737.81   156.8
 1097.57  156.23 1371.23  160.13 1475.98  156.35 1481.96  155.35 1499.92  147.25
 1518.83 142.3171554.886 142.2631660.065 142.306 1663.73  144.35 1676.72  146.82
 1745.62     149 1797.47   154.5 1872.26   156.1 1884.22  161.63 1895.19  162.87
 1900.18  165.21 1907.16  162.22 1926.11  161.63 1978.96  164.81 2017.84  163.42
 2123.51  165.28 2162.39  170.62 2222.21  174.02 2267.07  175.72 2317.91  175.08
#Mann= 3 , 0 , 0
       0     .12       0 1518.83    .035       0 1663.73     .12       0
Bank Sta=1518.83,1663.73
XS Rating Curve= 0 ,0
Exp/Cntr=0.3,0.1

Type RM Length L Ch R = 1 ,122.4162,604.52,574.75,568.14
BEGIN DESCRIPTION:
E36 (SEM 2016)
END DESCRIPTION:
XS GIS Cut Line= 6
     533634.1548    5403673.7426     533996.2002     5403176.955
     534064.3351    5402581.0789     534137.6282    5402503.1736
     534460.8021    5402159.6619     534840.1703    5401756.4189
#Sta/Elev= 30
       0  186.42  170.92  184.14  339.84  172.56  443.79  167.53  746.66  156.99
  939.58  152.79 1214.47  153.74 1431.42  152.53 1479.42  150.63 1507.41  152.58
 1558.41  152.42 1578.41   146.1  1595.4  144.251598.605  141.341628.516 139.333
 1672.31  143.15 1679.29  144.82 1712.23  146.04 1825.06   147.6 1887.02  157.03
 1931.99  157.99 1941.98  159.84 1969.97  160.79 2020.93  168.92 2084.89  170.74
 2095.89  173.05 2263.79  173.31 2283.78  170.56 2315.76  171.23 2346.74  169.39
#Mann= 3 , 0 , 0
       0     .12       01598.605    .035       0 1672.31     .12       0
Bank Sta=1598.605,1672.31
XS Rating Curve= 0 ,0
Exp/Cntr=0.3,0.1

Type RM Length L Ch R = 1 ,121.8414,339.5,326.96,323.17
XS GIS Cut Line= 6
     533786.2744    5403837.6298     534351.4758    5403099.0873
     534675.5884    5402749.0947     534825.7921    5402586.8972
     535036.3437    5402359.5329     535521.1549    5401819.8444
#Sta/Elev= 30
       0  190.43     179   187.2     532  165.36  940.96  154.42 1076.56  147.73
 1109.47  148.24 1118.44  149.98 1195.32  150.73 1291.18  149.39 1307.15  148.47
 1326.13     1431329.318 141.6781400.997 141.6421492.582 141.697 1495.63  143.28
 1508.57  149.19 1515.54  150.15  1595.2  148.87 1639.06  149.73 1654.05  152.54
 1760.01  152.65 1843.98   157.8 1890.96  157.96 1940.94  163.72 2043.87  167.26
 2212.74  167.47 2224.74  166.02 2352.64  164.84 2454.57  168.42 2663.41  168.29
#Mann= 3 , 0 , 0
       0     .12       0 1326.13    .035       0 1495.63     .12       0
Bank Sta=1326.13,1495.63
XS Rating Curve= 0 ,0
Exp/Cntr=0.3,0.1

Type RM Length L Ch R = 1 ,121.5145,510.63,436.62,421.87
XS GIS Cut Line= 6
     534552.3254    5404000.0554     534761.8651    5403242.2098
     534798.9354    5403108.1363     535012.9942    5402846.0645
     535274.1189    5402617.0239     535380.6256    5402414.7812
#Sta/Elev= 30
       0  180.26  201.82  167.78  278.75  166.31  340.69  167.94  403.63  166.14
  454.58  161.37  478.56  161.55  533.51  158.16   908.5  147.38  975.07  143.35
  981.03  142.96 982.801 141.658 1153.16 141.639 1165.12  143.55    1200  146.05
 1214.95  150.89 1353.61  149.01 1376.56  152.75 1399.52  154.42 1452.42  155.87
 1480.37  161.13 1497.33  161.03 1533.26  156.92 1550.23  157.07 1608.12  161.97
 1625.09  161.14 1695.96  165.32 1754.84  173.05 1806.75  174.26 1839.68  172.94
#Mann= 3 , 0 , 0
       0     .12       0  975.07    .035       0 1165.12     .12       0
Bank Sta=975.07,1165.12
XS Rating Curve= 0 ,0
Exp/Cntr=0.3,0.1

Type RM Length L Ch R = 1 ,121.0779,586.92,585.54,574.22
XS GIS Cut Line= 6
     535226.5108    5404275.0156      535241.194    5403923.7687
     535289.0529    5403236.9187      535299.743    5403083.4973
     535311.2315    5403050.6979     535513.5933    5402515.5628
#Sta/Elev= 30
       0  168.62   45.94  165.93  201.74   166.1  231.71  167.69  290.63  165.95
  483.46  167.09  532.43  165.33  751.27  164.77   862.2  161.81  937.14  163.95
 1039.07  160.42 1062.02   147.7    1070   145.2 1117.88  142.691119.606 141.496
1248.716 141.465 1256.57  143.07 1376.39  155.69 1424.31  156.85 1451.27   160.9
 1465.25  165.66 1477.23   164.8 1502.19  157.66 1507.18  158.83 1517.17  157.31
 1565.09  156.95 1659.94  165.55 1708.87  164.32 1736.82  168.65 1800.72  169.97
#Mann= 3 , 0 , 0
       0     .12       0 1117.88    .035       0 1256.57     .12       0
Bank Sta=1117.88,1256.57
XS Rating Curve= 0 ,0
Exp/Cntr=0.3,0.1

Type RM Length L Ch R = 1 ,120.4923,772.66,736.03,708.52
XS GIS Cut Line= 6
     535848.9593     5404253.562     535856.4625    5403936.2585
     535860.9884    5403310.9812     535861.5221    5403237.2468
      535862.131    5403153.1104     535867.3515     5402462.492
#Sta/Elev= 30
       0  176.86  148.72  178.38  204.61  175.88  362.34  175.81   399.3  178.18
  440.25  173.59  570.11  176.29  639.03     170  690.97  167.86  705.95   168.1
  722.93   171.9  744.91  174.05  791.86  172.99  824.82  169.79  864.77  170.63
  873.76  169.64  914.72  158.66   934.7  151.56  946.67  144.26  957.94 141.802
 1026.51 140.502 1081.07 141.802 1107.56  143.12 1150.53  151.65 1242.48   158.6
 1377.41  155.68 1519.33  163.49 1703.23  164.91  1758.2  168.99 1791.18  167.87
#Mann= 3 , 0 , 0
       0     .12       0  957.94    .035       0 1081.07     .12       0
Bank Sta=957.94,1081.07
XS Rating Curve= 0 ,0
Exp/Cntr=0.3,0.1

Type RM Length L Ch R = 1 ,119.7563,652.27,599.9,552.88
BEGIN DESCRIPTION:
E35 (SEM 2016)
END DESCRIPTION:
XS GIS Cut Line= 5
     537019.7128    5404041.3418     536623.6031    5403204.2395
     536582.5958    5403117.5784     536486.2617    5402913.9953
     535996.7578    5401879.5279
#Sta/Elev= 30
       0  213.08   22.98  215.13   64.94  212.08   66.93  209.32  106.89  206.99
  125.88  201.35   201.8  198.66  340.66   183.1  501.51  172.39  790.23  160.27
  872.15  149.79  938.08   148.9  955.06  141.61  972.04   140.41000.847 136.342
 1077.31   139.9 1110.67  144.34 1137.57   154.9 1478.08  152.57 1546.05  161.85
    1640  155.12 1701.97  157.55 1733.95  151.94 1971.83  151.71 2051.79  156.55
 2104.76  154.42 2171.73  159.53  2230.7  171.69 2308.66  171.08 2391.62  177.85
#Mann= 3 , 0 , 0
       0     .12       0  972.04    .035       0 1077.31     .12       0
Bank Sta=972.04,1077.31
XS Rating Curve= 0 ,0
Exp/Cntr=0.3,0.1

Type RM Length L Ch R = 1 ,119.1564,743.23,788.29,842.46
XS GIS Cut Line= 6
      537455.139    5403414.9229     537356.4462    5402953.3491
     537100.0565    5402799.7469     536950.1532    5402709.9404
     536928.5618     5402663.122     536530.3932    5401799.7467
#Sta/Elev= 30
       0  194.66  210.56  181.75  244.49  176.63  336.29  173.44  383.19  175.12
  400.16  171.08  502.99  160.75  583.96  159.11  623.94  161.54  645.93  156.52
   730.9  151.67  739.89  147.68  757.89  148.02  788.66  139.79 883.784 137.361
  921.47 137.465  962.48  143.44  986.28  153.05 1048.17  150.77 1084.16  153.57
 1132.15  150.51 1296.11  154.87  1352.1  170.55 1544.05  169.68 1604.03  173.71
 1651.02  172.68    1731  182.92 1814.98  185.41 1908.96  195.08 1947.95  194.14
#Mann= 3 , 0 , 0
       0     .12       0  788.66    .035       0  921.47     .12       0
Bank Sta=788.66,921.47
XS Rating Curve= 0 ,0
Exp/Cntr=0.3,0.1

Type RM Length L Ch R = 1 ,118.3681,240.68,238.12,238.92
XS GIS Cut Line= 3
     537788.0069     5403307.416      537741.781    5402604.3679
     537436.5626    5401448.9923
#Sta/Elev= 30
       0  185.03  243.85  174.04  297.82  166.01  343.79  162.06  531.67  156.68
  587.64  150.69   641.6  150.53  660.59  153.59  720.55  154.26  740.53  145.43
  747.53  143.86   778.5  142.02  954.36  139.53  972.88 135.7771001.852 135.729
 1094.25  136.68 1124.22  142.22  1146.2  152.68 1171.18   167.7 1194.17  172.33
 1241.13  172.06 1255.12  169.16  1271.1   171.6 1385.01  177.04 1451.96  175.79
 1582.85  176.94 1605.83  181.52 1804.67  189.04 1862.62  185.12 1899.59  185.18
#Mann= 3 , 0 , 0
       0     .12       0  972.88    .035       0 1094.25     .12       0
Bank Sta=972.88,1094.25
XS Rating Curve= 0 ,0
Exp/Cntr=0.3,0.1

Type RM Length L Ch R = 1 ,118.1300,354.68,394.02,459.66
BEGIN DESCRIPTION:
E34 (SEM 2016)
END DESCRIPTION:
XS GIS Cut Line= 4
     537913.4622    5403278.5398     537915.5012    5402317.9797
     537848.4943     5402102.515     537965.5614    5401322.8757
#Sta/Elev= 30
       0  181.46   35.98  181.14   79.96  175.83  192.91  171.94  272.88  173.18
  352.84  161.81  472.79   158.4  552.75  150.01  627.71  149.27  730.67  143.42
  982.03   139.1  987.52  137.83 989.738 134.6621052.836 133.761 1114.31  135.96
 1144.27  142.29 1157.24  148.64 1231.16  155.87 1267.13   166.6  1309.1  171.58
 1352.06  173.37 1380.04  180.82 1399.03  180.56 1445.99  185.89 1661.81   185.7
 1693.79  190.69 1727.76  190.76 1758.73  194.06 1812.69  192.83 1974.56  201.61
#Mann= 3 , 0 , 0
       0     .12       0 989.738    .035       0 1114.31     .12       0
Bank Sta=989.738,1114.31
XS Rating Curve= 0 ,0
Exp/Cntr=0.3,0.1

Type RM Length L Ch R = 1 ,117.7360,1127.18,1115.18,1111.76
XS GIS Cut Line= 3
     538024.0447    5403318.0837     538125.7692    5402649.1274
      538617.848    5401532.2877
#Sta/Elev= 30
       0  182.78   50.97  182.18  107.94   177.8  177.91  181.51  212.89  178.11
   374.8  174.35  481.75  165.24  600.68  150.86  708.63  150.17  734.62  153.61
  758.61  144.48   769.6  143.16  892.55   141.5 937.786 134.721 948.293 134.637
 1050.55 134.697 1054.48  136.35 1099.46  139.24 1172.42   153.2 1204.41  160.75
  1225.4  170.62 1239.39  173.05 1261.38  180.39 1299.36  184.68 1497.27  183.44
 1533.25   186.3 1655.19  184.34 1722.16  189.69 1742.15  193.01 1897.08  196.54
#Mann= 3 , 0 , 0
       0     .12       0 937.786    .035       0 1054.48     .12       0
Bank Sta=937.786,1054.48
XS Rating Curve= 0 ,0
Exp/Cntr=0.3,0.1

Type RM Length L Ch R = 1 ,116.6208,638.24,668.89,689.51
BEGIN DESCRIPTION:
E33 (SEM 2016)
END DESCRIPTION:
XS GIS Cut Line= 5
      538755.331    5403644.5839      539021.716    5403215.8555
     539201.5247    5403011.6316       539278.44    5402762.5032
     539866.5513     5401856.146
#Sta/Elev= 30
       0  185.19  150.92  179.49  170.91  177.35   394.8  171.11  660.24  154.56
  738.98  146.36  816.81   146.6  859.77  138.89  869.76  134.67 871.295 132.691
 979.709 131.2431015.152 131.984  1021.6  133.83  1024.6  135.26 1073.56  138.78
 1110.55  147.76 1152.52  154.52 1165.52  159.33 1182.51  158.75 1280.46  167.76
  1383.4  172.29 1465.36  171.31 1479.35  171.96 1489.35  174.44 1624.28  179.82
 1722.22  188.03 1964.09  194.44 2044.05  198.03 2061.05  200.62 2118.02  204.55
#Mann= 3 , 0 , 0
       0     .12       0 871.295    .035       0  1021.6     .12       0
Bank Sta=871.295,1021.6
XS Rating Curve= 0 ,0
Exp/Cntr=0.3,0.1

Type RM Length L Ch R = 1 ,115.9519,1338.41,1323.34,1310.4
XS GIS Cut Line= 2
     539310.9367    5403943.4952     540515.0906    5402168.9735
#Sta/Elev= 30
       0  188.13   47.99  185.33  195.95   182.1  395.91  170.75  503.88  160.23
  621.86  146.08  645.85  141.12  696.84     140  739.83   141.8  825.81  141.77
  850.81  140.13   873.8  134.15  892.34 133.146  957.79 131.146 1011.77 132.626
 1026.77  136.55 1123.75  145.02 1218.72  148.44 1277.71  154.89 1337.69  156.75
 1385.68  164.58 1472.66  165.06 1595.63  174.69 1666.61  177.33 1787.58   178.1
 1818.57  181.96 1936.54   185.6 1953.54  188.06 2028.52  191.99 2144.49  193.56
#Mann= 3 , 0 , 0
       0     .12       0  892.34    .035       0 1011.77     .12       0
Bank Sta=892.34,1011.77
XS Rating Curve= 0 ,0
Exp/Cntr=0.3,0.1

Type RM Length L Ch R = 1 ,114.6285,1781.96,1782.74,1777.07
BEGIN DESCRIPTION:
E32 (SEM 2016)
END DESCRIPTION:
XS GIS Cut Line= 3
     540338.6514    5404582.5478     540896.6122    5403993.0967
     541471.9812    5402722.4448
#Sta/Elev= 30
       0  187.69   228.9  174.02  254.89  171.74  277.88  166.83  564.75  151.66
   692.7  142.71  766.66  140.29  803.65  136.01  847.49  135.43  868.64  133.45
 870.591 131.144 912.063 129.418 992.822 131.422  998.62  134.98 1033.62  140.09
 1084.61  143.91 1133.61  151.11  1155.6   151.3  1205.6  157.07 1260.59  158.35
 1309.59  161.89 1380.58  160.66 1720.54  164.71 1765.54  163.05 1902.52  168.79
 2000.51  170.57  2098.5  177.75  2107.5  179.92  2147.5  179.75 2206.49  183.32
#Mann= 3 , 0 , 0
       0     .12       0 870.591    .035       0  998.62     .12       0
Bank Sta=870.591,998.62
XS Rating Curve= 0 ,0
Exp/Cntr=0.3,0.1

Type RM Length L Ch R = 1 ,112.8458,1633.09,1639.21,1638.27
BEGIN DESCRIPTION:
E31 (SEM 2016)
END DESCRIPTION:
XS GIS Cut Line= 5
     541622.4561    5405960.9932     542154.4075    5405276.2596
     542246.2378     5405066.233     542301.3958    5404912.5037
     542995.9474    5404184.4592
#Sta/Elev= 30
       0  227.04  124.87  221.29  223.76  208.93  435.54  194.06  464.51  195.88
  484.49  189.92  615.35  185.38  705.25  176.07  778.18  176.94  837.11  170.27
   951.8  167.74  998.64  144.311037.426 130.8811069.952 128.8751170.041  130.99
 1178.97  135.12 1264.63   150.7  1305.6  162.95 1334.58  166.98 1412.52  162.77
 1597.38  162.01 1660.33  152.95 1783.24  148.82 1843.19  148.68 1859.18  153.44
 1918.14  160.61 2007.07  162.65 2058.03  167.57 2139.97  167.93 2265.87  159.09
#Mann= 3 , 0 , 0
       0     .12       01037.426    .035       01170.041     .12       0
Bank Sta=1037.426,1170.041
XS Rating Curve= 0 ,0
Exp/Cntr=0.3,0.1

Type RM Length L Ch R = 1 ,111.2066,968.71,946.26,942.59
XS GIS Cut Line= 3
     543122.0861    5406823.4679     543655.0429    5405882.3909
     544202.4767    5404420.4283
#Sta/Elev= 30
       0  204.57   218.9  191.68  305.86  180.27  513.77  162.12  562.75  155.66
  784.65  144.48 1040.54  145.51 1054.53  138.46 1076.66  131.541162.176 131.053
 1227.44  131.55 1279.41  137.64 1403.34  140.64 1458.31  147.69 1533.26   150.9
 1578.24  157.42 1665.19  156.85 1692.17  154.19 1756.14  154.23 1792.12  156.57
 1848.09  151.55 1910.05  153.25 2072.96  149.15 2236.86  157.91 2307.82  163.79
 2465.72  163.52 2550.67  167.12 2562.67  165.66 2576.66  168.25 2642.62  170.22
#Mann= 3 , 0 , 0
       0     .12       0 1076.66    .035       0 1227.44     .12       0
Bank Sta=1076.66,1227.44
XS Rating Curve= 0 ,0
Exp/Cntr=0.3,0.1

Type RM Length L Ch R = 1 ,110.2603,1132.18,1175.64,1233.62
BEGIN DESCRIPTION:
E30 (SEM 2016)
END DESCRIPTION:
XS GIS Cut Line= 6
     543888.3727     5407326.105     544518.0009    5406391.0309
     544549.4521    5406330.1575     544515.7532    5406237.3407
     544514.7692    5406057.0446     545327.0652    5405097.5456
#Sta/Elev= 30
       0  192.64   159.9  178.63  215.87  177.54  438.73  162.84  677.57  160.68
  774.51  151.16  856.46  148.37   950.4  148.76 1017.36   153.1 1065.33  146.78
 1223.74  141.05    1257  129.881365.895  127.72 1414.25  130.37 1527.81  134.77
 1552.79  143.38 1578.78  146.42 1606.76  146.66 1634.74  135.47 1661.72  136.03
 1723.67  146.58 1804.62  146.91 1862.58   154.5 1987.49  155.92 2007.47  161.46
 2050.44  166.04 2249.31  177.41 2394.21  174.67 2597.07  186.83 2731.97  185.28
#Mann= 3 , 0 , 0
       0     .12       0    1257    .035       0 1414.25     .12       0
Bank Sta=1257,1414.25
XS Rating Curve= 0 ,0
Exp/Cntr=0.3,0.1

Type RM Length L Ch R = 1 ,109.0847,1038.86,996.34,970.72
XS GIS Cut Line= 2
      544574.635    5408345.1461     546255.7539    5405628.7522
#Sta/Elev= 30
       0   186.4      33  186.04   34.99  183.34   96.99  179.23  135.98  181.18
  335.95  171.76  422.94  172.22  935.87  150.43  1383.8   140.1 1532.78  140.86
 1619.76  138.16 1757.28 129.534 1820.36 127.744 1877.72 129.674 1894.72  141.79
 1899.72  143.22 2241.65  144.99 2320.63  152.53 2542.58  158.82 2677.55  171.35
 2767.52   175.4  2857.5  187.25 2934.48  203.61 2963.48  207.46 3043.46  235.79
 3061.45  246.57 3108.44  249.85 3136.44  259.06 3163.43  273.93 3194.42  279.68
#Mann= 3 , 0 , 0
       0     .12       0 1757.28    .035       0 1877.72     .12       0
Bank Sta=1757.28,1877.72
XS Rating Curve= 0 ,0
Exp/Cntr=0.3,0.1

Type RM Length L Ch R = 1 ,108.0884,1472.46,1471.09,1474.86
BEGIN DESCRIPTION:
E29 (SEM 2016)
END DESCRIPTION:
XS GIS Cut Line= 5
     546333.6993    5408244.5183     546435.9397    5407234.9086
     546453.8595    5407120.1978      546509.894    5406921.6061
     546966.8596    5405444.2896
#Sta/Elev= 30
       0   183.2  255.94  184.54  332.93  181.19  365.92  176.97  508.89  173.33
  555.88  166.65  596.87  167.95  654.85   159.2  848.81  145.56   894.8  138.71
 1008.77  129.781065.053 124.544    1114  128.45 1162.77  137.63 1178.72  144.26
 1253.48  141.65 1471.15  141.78 1499.14  147.03 1568.11  145.58  1595.1  149.46
 1714.05  152.61    1828  164.15 1908.97  176.11 2050.91  208.73 2138.88  224.75
 2236.84   236.8 2515.74   247.4  2634.7  241.83 2823.63   241.8  2883.6  244.36
#Mann= 3 , 0 , 0
       0     .12       0 1008.77    .035       0    1114     .12       0
Bank Sta=1008.77,1114
XS Rating Curve= 0 ,0
Exp/Cntr=0.3,0.1

Type RM Length L Ch R = 1 ,106.6173,1956.56,1954.42,1973.2
BEGIN DESCRIPTION:
E28 (SEM 2016)
END DESCRIPTION:
XS GIS Cut Line= 2
     547655.8825    5408699.5296     548236.2092     5405539.685
#Sta/Elev= 30
       0  206.15  181.98  197.65  199.98  191.71  550.95  165.03  656.94  161.03
  684.93  155.63  766.92  156.66  919.91   149.7 1077.89  137.39 1198.89   132.4
 1210.88  134.65 1221.88  130.26 1253.88  127.331357.594 124.4641398.168 126.067
 1447.87  139.36 1540.87  146.92 1644.86   149.6 1737.86  159.71 1838.85  165.22
 1910.85  164.76 2063.84  178.55 2147.83  178.74 2195.82  185.86 2286.81  182.86
  2420.8  186.54 2597.78  201.66 2785.76  206.47 2973.74  199.79 3212.72  205.95
#Mann= 3 , 0 , 0
       0     .12       0 1253.88    .035       01398.168     .12       0
Bank Sta=1253.88,1398.168
XS Rating Curve= 0 ,0
Exp/Cntr=0.3,0.1

Type RM Length L Ch R = 1 ,104.6629,381.74,383.17,410.51
BEGIN DESCRIPTION:
E27 (SEM 2016)
END DESCRIPTION:
XS GIS Cut Line= 4
     549617.3781    5408956.9241     549800.8356    5407793.9656
     549867.5497    5407443.6106     549619.4807    5405404.6342
#Sta/Elev= 30
       0  202.08   180.9   191.2  317.82  170.99  430.76  160.61  652.63  154.01
  688.61   155.3   874.5  141.52  996.43  135.96 1073.39  136.45 1102.37     132
  1213.3  132.03 1243.27  126.891427.933 124.1871458.398 125.598 1483.03  140.05
 1706.89  140.28 1759.87  137.16 2001.75  135.69 2172.67  143.59  2316.6  139.11
 2347.58  140.37 2467.52  156.57 2593.46  144.81 2707.41  149.87 2789.36  157.71
 3143.19   179.1 3452.04  187.38 3461.04  187.76 3464.04  190.63 3587.97   191.5
#Mann= 3 , 0 , 0
       0     .12       0 1243.27    .035       01458.398     .12       0
Bank Sta=1243.27,1458.398
XS Rating Curve= 0 ,0
Exp/Cntr=0.3,0.1

Type RM Length L Ch R = 1 ,104.2797,330.77,334.7,388.73
XS GIS Cut Line= 3
     549808.6149    5409016.4732      550193.652    5407788.8907
     550485.1929    5406077.4632
#Sta/Elev= 30
       0  198.01  171.94  186.01  370.87  164.75  511.82  158.62  527.82  153.72
  725.75  149.21  803.72  139.12 1167.59  136.88 1230.57  126.621253.718 125.453
 1301.54  127.48 1488.45  128.24 1632.37  127.38 1648.37  130.85 1905.23  133.62
  1965.2  133.45 1979.19  128.64 2251.05  129.24 2266.05  132.98 2337.01  130.33
    2364  131.53 2376.99  137.27 2409.97  138.09 2560.89  134.44 2608.87  144.81
 2621.86  154.24 2763.79     145 2856.74  153.93 2978.68  154.68 3022.65  158.84
#Mann= 5 ,-1 , 0
       0     .12       0 1230.57    .035       0 1301.54     .12       0
 1488.45    .035       0 1632.37     .12       0
Bank Sta=1230.57,1632.37
XS Rating Curve= 0 ,0
Exp/Cntr=0.3,0.1

Type RM Length L Ch R = 1 ,103.9450,347.77,362,388.94
XS GIS Cut Line= 4
     549950.6288    5409107.3847     550464.4224    5407966.8424
     550610.4564    5407565.2158     551130.9313    5406612.8083
#Sta/Elev= 30
       0  198.93      72  193.64      87  188.21  100.99  190.72  245.99  173.52
  385.98  161.54  582.97  150.35  610.97  144.77  703.96  139.21 1016.94  138.79
 1105.93  141.68 1305.84  136.35 1326.81  128.96 1370.34 125.909 1558.46  127.96
 1651.32   135.9 1754.23  127.38 1942.12  129.16  1968.1  134.62 2127.01  131.96
 2154.99   135.9 2233.94  133.99 2275.92  142.37 2375.86  150.03 2480.79   143.3
 2511.77  149.02 2554.75  150.07 2595.72  155.48 2650.69  168.15 2763.62   203.9
#Mann= 3 , 0 , 0
       0     .12       0 1370.34    .035       0 1558.46     .12       0
Bank Sta=1370.34,1558.46
XS Rating Curve= 0 ,0
Exp/Cntr=0.3,0.1

Type RM Length L Ch R = 1 ,103.5830,1112.46,1129.1,1151.32
BEGIN DESCRIPTION:
Noel Pauls Brook - E26 (SEM 2016)
END DESCRIPTION:
XS GIS Cut Line= 4
     550181.3612    5409195.5247     550667.0741    5408269.4761
     551000.5337    5407682.3974     551712.5564    5407197.5705
#Sta/Elev= 30
       0  191.64   69.98  181.05  114.97  179.45  214.94  167.51  257.93  166.72
  289.92  161.79   330.9  160.94   362.9  154.62  570.84  139.86  896.74  138.78
  944.73  145.09  998.71  145.82 1194.52   137.1 1306.38  138.22 1313.37  137.11
 1324.36  129.761325.299 125.0951353.652   123.5 1485.16  126.33  1833.8  135.41
 1872.77  138.69 2045.65  134.15 2220.53  150.77  2258.5  146.95 2349.43  148.93
 2462.35     162 2496.33  179.76  2532.3  185.21 2567.28  185.64 2582.27  189.37
#Mann= 3 , 0 , 0
       0     .12       01325.299    .035       0 1485.16     .12       0
Bank Sta=1325.299,1485.16
XS Rating Curve= 0 ,0
Exp/Cntr=0.3,0.1

Type RM Length L Ch R = 1 ,102.4539,446.11,446.73,454.81
XS GIS Cut Line= 2
     550764.5705    5409706.2411     552602.3674    5407707.2283
#Sta/Elev= 30
       0  178.05   33.99   170.9  126.97  166.86  208.96  155.83  373.92  144.18
  565.88   137.3  870.82  139.75  899.82   135.1 1080.78  133.79 1120.77  129.49
 1133.77  133.27 1165.76  132.85 1197.64  125.681361.442 124.278 1475.18 126.338
 1483.68  131.32 1704.63  143.71 1872.59  139.27 1897.59  144.55 2067.55  154.58
 2153.53  166.08 2311.49   171.6 2369.48  177.59 2377.48  183.19 2407.47  182.26
 2458.46  188.14 2532.44  187.54 2591.43  197.55 2602.43  202.83  2715.4  213.24
#Mann= 3 , 0 , 0
       0     .12       0 1197.64    .035       0 1475.18     .12       0
Bank Sta=1197.64,1475.18
XS Rating Curve= 0 ,0
Exp/Cntr=0.3,0.1

Type RM Length L Ch R = 1 ,102.0072,467.27,460.36,459.14
XS GIS Cut Line= 2
     551052.8398    5409993.6098     552983.5166    5408012.7473
#Sta/Elev= 30
       0  174.54  140.95  156.59  283.91  145.62  528.83  141.85  677.78  133.52
  828.72  137.72 1177.61  137.69  1210.6 125.0651221.752 124.967 1283.58  126.53
 1402.54  125.66 1549.49  125.68 1568.49  136.38 1871.39  139.12 1982.36   144.4
  2202.3  167.97 2309.27  171.65 2476.23  192.24 2495.22  196.79 2504.22  202.05
 2565.21  204.52  2569.2  208.25  2592.2  208.25  2597.2  211.88 2647.18   215.4
 2651.18  219.78 2753.16  228.02 2759.16  229.92 2761.15  233.33 2766.15  233.33
#Mann= 5 ,-1 , 0
       0     .12       0  1210.6    .035       0 1283.58     .12       0
 1402.54    .035       0 1549.49     .12       0
Bank Sta=1210.6,1549.49
XS Rating Curve= 0 ,0
Exp/Cntr=0.3,0.1

Type RM Length L Ch R = 1 ,101.5468,909.18,894.07,898.57
BEGIN DESCRIPTION:
E25 (SEM 2016)
END DESCRIPTION:
XS GIS Cut Line= 2
     551420.3214    5410289.3998     553342.8148    5408287.2667
#Sta/Elev= 30
       0   170.5  129.99  157.74  509.94  141.09  541.94  135.68 1197.87   136.1
 1243.86  124.881340.551 123.375 1480.84  125.12 1514.84  134.44 1544.83  132.21
 1680.82  138.76  1856.8  135.95 2219.76  162.96 2280.75  173.99 2363.75  179.66
 2369.74  183.26 2397.74  181.32 2422.74  188.91 2458.74  187.66 2484.74  197.17
 2501.73  197.68 2522.73  205.09 2552.73  206.86 2561.73  211.89 2587.73   215.5
 2636.72   215.5 2640.72   219.2 2691.72  222.84 2694.71  227.05  2775.7  232.21
#Mann= 3 , 0 , 0
       0     .12       0 1243.86    .035       0 1480.84     .12       0
Bank Sta=1243.86,1480.84
XS Rating Curve= 0 ,0
Exp/Cntr=0.3,0.1

Type RM Length L Ch R = 1 ,100.6527,1731.24,1744.38,1770.48
XS GIS Cut Line= 3
     552146.8385    5411129.6135     553138.4007    5409754.3654
     554204.5836      5408820.28
#Sta/Elev= 30
       0  164.11   97.97  155.59  184.94  154.52  355.88  144.18  559.81  142.66
  795.73  134.28 1017.65  131.06  1491.5  135.33  1504.5  134.461524.111 123.708
1625.879 123.6961754.732 123.746  1779.4  126.96 1847.38  143.65 1974.33  153.42
 2123.27  169.32 2180.25  165.98 2222.23  169.96  2292.2  168.84 2359.18  174.04
 2416.15  173.55 2491.12  179.97 2530.11  179.18 2648.06  186.03 2665.05  189.71
 2706.03  191.18 2732.02   198.5 2844.98  205.28 3008.91   206.4 3112.87  202.61
#Mann= 3 , 0 , 0
       0     .12       01524.111    .035       01754.732     .12       0
Bank Sta=1524.111,1754.732
XS Rating Curve= 0 ,0
Exp/Cntr=0.3,0.1

Type RM Length L Ch R = 1 ,98.9083 ,596.7,523.2,496.56
BEGIN DESCRIPTION:
DS of 02YO011 ER below NP Brook - E24 (SEM 2016)
END DESCRIPTION:
XS GIS Cut Line= 5
     553759.6838    5412399.4191     554178.1701    5411302.7808
     554221.8514    5411134.8619     554386.8006    5410950.5432
     554801.0484    5410113.1202
#Sta/Elev= 30
       0  157.15  118.98  157.11  301.94  152.82  702.86  137.46  780.85  138.08
  829.84  134.34  939.82  133.97  969.81  137.16 1102.79  136.74 1211.67  132.26
 1222.64   135.2 1232.61  134.36 1241.58  130.47 1315.37  126.97 1333.56  123.78
1358.799  120.92 1591.63  123.83 1635.59  128.24 1736.51  128.61 1962.34  137.05
 2021.29  141.94 2065.26     143 2117.22  151.29  2144.2   151.7 2192.17  158.09
 2239.13   159.5 2298.09  168.73 2351.05  170.25 2400.02   167.5 2528.92  176.89
#Mann= 3 , 0 , 0
       0     .12       0 1333.56    .035       0 1591.63     .12       0
Bank Sta=1333.56,1591.63
XS Rating Curve= 0 ,0
Exp/Cntr=0.3,0.1

Type RM Length L Ch R = 1 ,98.3851 ,801.76,784.8,779.52
XS GIS Cut Line= 2
     554101.4056    5412484.3301     555320.9233    5410189.3732
#Sta/Elev= 30
       0  151.89  156.99  153.47  394.98  149.59  592.97  135.37  701.96  130.56
  884.95  130.82 1140.94   137.5 1235.93  135.92 1284.93  140.38 1314.92  137.22
 1339.92  125.78 1478.01 124.529  1540.8 119.959  1604.9 124.019  1626.9  128.97
 1748.89  140.11 1792.89  145.07 1819.88  151.16 1904.88  159.18 1914.88  163.15
 1973.87  170.52 2030.87   157.5 2045.87  156.62 2158.87  159.24 2229.87  168.61
 2264.87   171.2 2484.87  181.81 2539.87  180.81 2585.87  174.16 2598.87  170.36
#Mann= 3 , 0 , 0
       0     .12       0 1478.01    .035       0  1604.9     .12       0
Bank Sta=1478.01,1604.9
XS Rating Curve= 0 ,0
Exp/Cntr=0.3,0.1

Type RM Length L Ch R = 1 ,97.6003 ,137.83,133.04,131.81
XS GIS Cut Line= 2
     554720.9829    5412682.9408     556094.5787     5410580.473
#Sta/Elev= 30
       0   149.6  159.96   147.1  570.86  129.09  746.82  128.56  857.79  130.87
  956.77  128.49  967.76  131.26  979.76  127.45 1049.74  129.43 1161.75  123.25
 1250.82  120.56 1334.24  123.25 1348.67  126.82 1363.67  134.44 1390.66  137.34
 1586.62  139.09  1654.6  142.04 1790.57  141.85 1853.56  147.58 1908.54  147.96
 1948.53  152.42 2262.46  160.85 2411.42  175.07 2413.42  178.16 2417.42  179.54
 2433.42  179.54 2436.42  182.92 2456.41  184.14 2458.41  187.27  2511.4  190.75
#Mann= 3 , 0 , 0
       0     .12       0 1161.75    .035       0 1334.24     .12       0
Bank Sta=1161.75,1334.24
XS Rating Curve= 0 ,0
Exp/Cntr=0.3,0.1

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
Type RM Length L Ch R = 1 ,96.5359 ,121.35,128.61,131.24
BEGIN DESCRIPTION:
E23 (SEM 2016)
END DESCRIPTION:
XS GIS Cut Line= 4
     555469.8749    5413161.3214     556238.4071    5412274.6128
     556446.8978    5411909.6474     557000.9595    5411014.8591
#Sta/Elev= 30
       0  148.35  149.92  151.93  220.89  144.76  271.86  147.66  571.71  133.24
  642.68  132.74  760.62  134.61  867.57  144.01  988.51  140.63 1087.46  132.58
 1227.33  135.65 1300.22  140.96 1365.11  126.34 1419.72 119.4921465.579 117.331
 1532.85  120.76 1626.73   147.2 1643.72  149.11 1725.68  148.04 1763.66  152.44
 1794.64  149.07 1831.62  150.92 1953.55  146.72  2059.5  154.81 2093.48  162.38
 2219.41  167.47 2359.34  183.38 2495.27  187.21 2543.25  192.81 2646.19  197.42
#Mann= 3 , 0 , 0
       0     .12       0 1419.72    .035       0 1532.85     .12       0
Bank Sta=1419.72,1532.85
XS Rating Curve= 0 ,0
Exp/Cntr=0.3,0.1

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
Type RM Length L Ch R = 1 ,96.0215 ,123.43,143.77,169.66
XS GIS Cut Line= 4
     555567.9158    5413295.1012     556303.2225    5412553.2616
      556671.028    5412450.3883     557744.2909    5411300.5327
#Sta/Elev= 30
       0  148.89  113.95  149.13  151.93  153.68  174.92  150.21  259.88  149.72
  390.82  141.47  500.77  139.51  593.72   133.6  610.71  135.86  625.71  131.17
  968.55  130.06  997.53  132.56 1018.52  129.66 1160.49  129.58 1224.48  134.03
 1331.46  126.87 1379.45  120.01 1426.81 119.617 1561.44  120.29 1642.44  134.82
 1701.44  139.33 1805.44  139.72 1921.44  146.59 2136.43  148.52 2337.43  158.43
 2387.43  165.14 2441.43  164.07 2509.43  171.83 2640.43  179.74 2999.43  187.28
#Mann= 3 , 0 , 0
       0     .12       0 1379.45    .035       0 1561.44     .12       0
Bank Sta=1379.45,1561.44
XS Rating Curve= 0 ,0
Exp/Cntr=0.3,0.1

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
Type RM Length L Ch R = 1 ,95.4464 ,190.23,135.95,113.68
BEGIN DESCRIPTION:
Red Indian Falls
END DESCRIPTION:
XS GIS Cut Line= 5
      555791.468    5413223.1929     556299.3981    5412899.7288
     556393.2222    5412845.9387      557310.269    5413041.6158
     558005.2837    5412888.2945
#Sta/Elev= 30
       0  153.71  164.78  145.91  210.71  141.54  300.59  140.92  327.56  137.76
  374.49   139.7  503.32  131.52  697.43   130.7  962.25  132.73  986.24  123.67
 1016.23  123.14 1042.23  118.77 1052.22  114.44 1067.22  114.89 1078.21  118.44
 1089.21  118.71 1096.21  115.57  1115.2  114.881170.494  111.491233.718   112.8
 1236.17  114.92 1248.17  116.21 1258.16  119.86 1295.15  121.87 1312.15  126.19
 1493.09   126.1 1809.98  132.52 1899.95  135.28 1922.94  140.37 2359.77  136.07
#Mann= 3 , 0 , 0
       0     .12       0  1115.2    .035       0 1236.17     .12       0
Bank Sta=1115.2,1236.17
XS Rating Curve= 0 ,0
Exp/Cntr=0.3,0.1

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
Type RM Length L Ch R = 1 ,94.9026 ,168.99,142.51,118.79
BEGIN DESCRIPTION:
E22 (SEM 2016)
END DESCRIPTION:
XS GIS Cut Line= 3
     555903.3233    5414018.7943     557105.7759    5413304.4824
     558149.2571    5412925.5934
#Sta/Elev= 30
       0  178.08  149.96  163.56  322.91  151.99   371.9  152.21  434.88  148.73
  478.87  142.38  499.86  142.22  526.86  138.28  667.82  132.54  681.82  133.87
  690.82  131.73   753.8  129.07  805.79  124.34  855.78  112.75  863.89  112.58
 1230.48 109.5611354.122 112.205 1355.65  115.04 1368.64  125.83 1386.64  126.59
 1652.44  127.52  1819.3     132 2018.15  133.86 2042.13  141.48 2053.12  141.45
  2072.1  136.41 2098.09  135.18 2155.04  136.92 2419.85  135.35 2508.78  140.03
#Mann= 3 , 0 , 0
       0     .12       0  863.89    .035       01354.122     .12       0
Bank Sta=863.89,1354.122
XS Rating Curve= 0 ,0
Exp/Cntr=0.3,0.1

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
Type RM Length L Ch R = 1 ,93.7625 ,137.08,146.91,159.07
BEGIN DESCRIPTION:
E21 (SEM 2016)
END DESCRIPTION:
XS GIS Cut Line= 4
     557156.0479     5415157.159     557860.0022    5414086.8477
     557855.4735     5413626.493     559040.6031    5413146.0574
#Sta/Elev= 30
       0  212.33   26.98  212.33   28.98  209.79   46.97  207.92   47.96  205.52
  342.75  170.61  525.62  155.97  570.58  146.02  695.49  143.24  778.43   136.8
  941.31  131.68 1102.19   131.1 1305.02  124.08 1312.01  123.741333.947 110.233
1378.023 110.155 1605.62  111.49 1703.49  124.84 1804.43  131.32 2393.32  134.09
 2518.29  141.84 2541.28  136.92 2619.27  135.87 2849.21  142.47 2888.21  146.72
 2937.19  138.38 2968.19  144.12 2986.18  144.82 3009.18  140.29 3020.18  142.23
#Mann= 3 , 0 , 0
       0     .12       01333.947    .035       0 1605.62     .12       0
Bank Sta=1333.947,1605.62
XS Rating Curve= 0 ,0
Exp/Cntr=0.3,0.1

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
Type RM Length L Ch R = 1 ,92.4404 ,117.01,124.5,132.94
BEGIN DESCRIPTION:
E20 (SEM 2016)
END DESCRIPTION:
XS GIS Cut Line= 3
      557492.581    5415516.0646     558660.5478    5414953.8789
      559819.038    5413697.0079
#Sta/Elev= 30
       0   212.4  151.91  203.55  154.91  199.61  235.86  190.48  412.75  175.85
  565.66  168.15   669.6  149.37   829.5  141.64  901.46  132.62 1074.36  119.58
 1286.23  119.66 1477.16  115.12 1493.15  110.151560.567 108.361  1708.3 108.879
 1709.07  112.14 1728.06  125.05 1778.04   123.2 1825.02  128.47 1932.98  123.57
 2089.92  127.59 2195.87  124.88 2395.77  130.84 2436.75  139.22 2461.74  136.35
  2544.7   140.1 2572.69   147.2 2863.56  142.67 2903.54  148.64 3005.49  148.97
#Mann= 3 , 0 , 0
       0     .12       0 1493.15    .035       0  1708.3     .12       0
Bank Sta=1493.15,1708.3
XS Rating Curve= 0 ,0
Exp/Cntr=0.3,0.1

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
Type RM Length L Ch R = 1 ,91.8179 ,420.96,355.52,291.8
XS GIS Cut Line= 4
     558039.5376    5415805.7839     559435.0019     5415131.463
     559579.0629    5414991.1417      560028.681    5414016.7805
#Sta/Elev= 30
       0  201.97  225.98  184.82  480.95  157.57  551.95  160.82  625.94     149
  748.93  141.75  876.92  129.78  928.91  118.82  1056.9  112.31 1134.89  114.16
 1181.09 109.0851224.629  109.06 1346.32 109.092 1366.86  124.96 1505.84  124.67
 1519.84  120.84 1543.84  120.25 1721.08  120.79 1824.89  125.82 2022.72  120.14
 2036.71  123.91 2151.62  122.24 2298.49  127.13 2442.37  127.61 2509.31  133.13
 2532.29  138.93 2568.26  133.77 2610.23  134.62  2641.2  140.21 2824.05   140.1
#Mann= 3 , 0 , 0
       0     .12       0 1181.09    .035       0 1346.32     .12       0
Bank Sta=1181.09,1346.32
XS Rating Curve= 0 ,0
Exp/Cntr=0.3,0.1

Type RM Length L Ch R = 1 ,91.4623 ,303.52,251.36,212.34
BEGIN DESCRIPTION:
E19 (SEM 2016)
END DESCRIPTION:
XS GIS Cut Line= 2
     558834.3882    5416435.7852     560253.7216    5414075.7224
#Sta/Elev= 30
       0  195.75      78  193.16     124  186.72     227  182.11     428  163.49
     575  154.29  706.99  137.34  809.99  130.05  905.99  117.99  947.99  109.34
1024.777 106.436 1133.99  109.38 1145.99  118.89 1167.99  118.47 1193.99  123.41
 1429.99  119.72 1714.98  124.21 1774.98   118.1 1912.98  122.15 1937.98  119.07
 1994.98  119.74 2074.98  128.72 2183.98  126.48 2239.98  129.44 2267.98  127.29
 2484.98  130.17 2516.98  135.09 2579.98  135.66 2629.98  140.17 2753.98  138.13
#Mann= 3 , 0 , 0
       0     .12       0  947.99    .035       0 1133.99     .12       0
Bank Sta=947.99,1133.99
XS Rating Curve= 0 ,0
Exp/Cntr=0.3,0.1

Type RM Length L Ch R = 1 ,91.2110 ,1131.72,1120.2,1130.16
XS GIS Cut Line= 3
     559566.2041    5416508.3709     559635.9532    5415259.6026
     560326.9877     5414080.171
#Sta/Elev= 30
       0  159.23  295.93  142.05  396.91  141.08   420.9  137.79  504.88  133.68
  543.88  129.42  567.87  128.24  583.87  129.83  596.86  126.08  712.84  118.23
  729.83  116.33  734.83  113.02  818.48 110.354  909.35 106.664  988.78 110.354
 1000.77  118.55 1042.76  120.44 1250.72  119.38 1354.72  123.32 1515.72   123.1
 1550.72  122.58 1577.72  117.17 1672.72  117.79 1832.72  119.82 1907.72  126.18
 1941.72  124.61 2344.72  130.41 2455.72   137.4 2487.72   133.5 2617.72  132.84
#Mann= 3 , 0 , 0
       0     .12       0  818.48    .035       0  988.78     .12       0
Bank Sta=818.48,988.78
XS Rating Curve= 0 ,0
Exp/Cntr=0.3,0.1

Type RM Length L Ch R = 1 ,90.0907 ,125.2,125.64,135.28
XS GIS Cut Line= 3
     560569.4322    5416541.1423     560705.8655    5415475.0354
     560743.0881    5413957.2947
#Sta/Elev= 30
       0  149.47      20  146.54  119.98  146.82  201.96  134.87  263.95  138.59
  310.94  128.91  349.93  130.49  375.93  125.72  469.91  120.72   531.9  122.89
  583.89  116.29  751.86  118.55  836.84  126.09  901.83  124.61  933.82  131.48
  974.81  130.67  1005.8   127.9  1030.8  109.86  1037.8  107.951178.618 106.445
 1220.71  107.53 1411.61  116.53 1567.53  127.98 1673.48  128.54 1704.46  134.95
 2243.18     136 2291.16  142.15 2443.09  143.05 2446.08  145.68 2593.01  149.01
#Mann= 3 , 0 , 0
       0     .12       0  1037.8    .035       0 1220.71     .12       0
Bank Sta=1037.8,1220.71
XS Rating Curve= 0 ,0
Exp/Cntr=0.3,0.1

Type RM Length L Ch R = 1 ,89.9651 ,130.8,162.48,192.3
BEGIN DESCRIPTION:
E18 (SEM 2016)
END DESCRIPTION:
XS GIS Cut Line= 2
     560662.7215    5416528.0841     561051.8143    5413976.6972
#Sta/Elev= 30
       0  143.32      92  141.26  131.99     135  182.99  132.22  209.99  133.41
  261.99   127.7  356.98  126.37  449.98  121.42  527.98  121.61  553.98  115.58
  585.97  114.81  764.97  119.12  800.97   123.6  896.96  125.29  932.96  129.88
  973.96  122.56 1027.96  120.98 1047.96  106.841103.852 104.029 1199.94  106.85
 1306.93  117.79 1525.91  126.13 1561.91  133.81  1652.9  132.32 1750.89  135.36
 2059.87  137.03 2110.87  141.78 2184.87  141.87 2369.87  148.35 2580.87  149.37
#Mann= 3 , 0 , 0
       0     .12       0 1047.96    .035       0 1199.94     .12       0
Bank Sta=1047.96,1199.94
XS Rating Curve= 0 ,0
Exp/Cntr=0.3,0.1

Type RM Length L Ch R = 1 ,89.8026 ,1217.88,1187.52,1165.32
XS GIS Cut Line= 3
     560756.4358    5416563.1777     560900.2033     5415608.496
     561729.4406    5414235.1136
#Sta/Elev= 30
       0  141.14  306.82  129.45   340.8  125.18  378.78  123.39  551.68  120.57
  579.67  115.25  595.66  114.53  764.56  117.08  779.55  119.33  825.53  119.22
  844.52  121.84  933.47  124.78  975.44  117.88 1023.42  115.09 1042.42  106.85
1050.695 106.2391188.907 106.251 1193.35  107.56 1203.35  109.87 1243.33  112.01
 1265.32  115.92 1443.25  121.99 1460.24  126.01 1755.11  130.25 1805.09  135.41
 1925.04  141.62 1971.02  138.61    2029  141.81 2490.77  146.67 2569.73   149.2
#Mann= 3 , 0 , 0
       0     .12       0 1042.42    .035       0 1193.35     .12       0
Bank Sta=1042.42,1193.35
XS Rating Curve= 0 ,0
Exp/Cntr=0.3,0.1

Type RM Length L Ch R = 1 ,88.6151 ,1054.24,1081.96,1119.36
BEGIN DESCRIPTION:
E17 (SEM 2016)
END DESCRIPTION:
XS GIS Cut Line= 4
     561463.5271    5417063.8699     561880.0633    5416369.7731
     562085.4953    5415835.4598     562636.1641    5414558.3531
#Sta/Elev= 30
       0  145.93   72.95  145.65  105.93     140   160.9  136.51  335.79  131.95
  398.75  134.45  556.65  126.37  686.56  127.44  720.54  130.69  739.53  126.53
   792.5  124.79  831.46  118.41  906.39  116.23  921.38  112.78  988.31  113.41
 1005.11  105.791034.612 103.488 1224.08  105.79 1234.07  110.46 1260.04   108.8
    1305  113.28 1381.92  130.63 1438.91   136.4 1573.89  130.52 1750.87  128.23
 1870.85  133.89 2277.78  143.65 2323.77   149.8 2448.75  155.29 2772.68   160.9
#Mann= 3 , 0 , 0
       0     .12       0 1005.11    .035       0 1224.08     .12       0
Bank Sta=1005.11,1224.08
XS Rating Curve= 0 ,0
Exp/Cntr=0.3,0.1

Type RM Length L Ch R = 1 ,87.5331 ,1263.46,1218.22,1177.28
XS GIS Cut Line= 3
     562350.6952     5417638.073     562916.2065    5416477.3041
     564123.2949    5415130.2685
#Sta/Elev= 30
       0  150.68   50.97  147.26   72.95  140.84   88.94  139.59  213.87  137.62
  293.82  139.87  354.78  132.81  525.67  128.08  683.57  119.51  864.46  119.01
 1011.37  115.22 1057.34  109.95 1296.19  109.52    1349  108.04 1362.18  105.25
1522.643 104.634 1531.16  106.12 1550.16  116.58 1601.15  133.23 1637.14   136.7
 1812.12  134.64 1961.09  138.94 2076.08  139.43 2265.04   146.1 2295.03  150.13
 2441.01  153.48    2473  157.76 2617.97  157.66  2982.9  170.05 3099.88   170.9
#Mann= 3 , 0 , 0
       0     .12       0 1362.18    .035       0 1531.16     .12       0
Bank Sta=1362.18,1531.16
XS Rating Curve= 0 ,0
Exp/Cntr=0.3,0.1
